--- bbc.prj (project) ---

Proj Title=bobong-ch
Current Plan=p01
Default Exp/Contr=.3,.1
SI Units
Geom File=g01
Flow File=f01
Plan File=p01
Y Axis Title=Elevation
X Axis Title(PF)=Main Channel Distance
X Axis Title(XS)=Station
BEGIN DESCRIPTION:
           BACK WATER COMPUTATION
      APPLICATION OF HEC-2 BY Samju Construction Engineering
      bobong-ch: 10,20,30,50,80 yr
END DESCRIPTION:
DSS Export Rating Curves= 0
DSS Export Rating Curve Sorted= 0
DSS Export Volume Flow Curves= 0
DXF OffsetX= 0
DXF OffsetY= 0
DXF ScaleX= 1
DXF ScaleY= 10

--- bbc.p01 (plan) ---

Plan Title=Imported Plan 01
Version=Version 3.0.1  Mar 2001
Short Identifier=Imported Pla
Geom File=g01
Flow File=f01
Subcritical Flow
K Sum by GR= 0
Std Step Tol= 0.003
Critical Tol= 0.003
Num of Std Step Trials= 20
Max Error Tol= 0.1
Flow Tol Ratio= 0.001
Split Flow NTrial= 30
Split Flow Tol= 0.02
Split Flow Ratio= 0.02
Log Output Level= 0
Friction Slope Method= 1
Unsteady Friction Slope Method= 2
Parabolic Critical Depth
Global Vel Dist= 0 , 0 , 0
Global Log Level= 0
CheckData=True
Encroach Param=-1 ,0,0, 0
Computation Interval=1HOUR
Output Interval=1HOUR
Run HTab= 0
Run UNet= 0
Run PostProcess= 0
UNET Theta= 1
UNET ZTol= 0.02
UNET ZSATol= 0.1
UNET MxIter= 20
UNET MaxInSteps= 20
UNET DtIC= 0
UNET DtMin= 0
UNET MaxCRTS= 20
UNET WFStab= 2
UNET SFStab= 1
UNET WFX= 1
UNET SFX= 1
UNET Convert EG Bridges=-1
UNET Use Existing IB Tables=-1
Instantaneous Interval=1HOUR
Write IC File= 0
Write Velocity= 0
Write Detailed= 0

--- bbc.f01 (steady flow) ---

Flow Title=Imported Flow 01
Version=Version 3.0.1  Mar 2001
Number of Profiles= 5
Profile Names=10yr,20yr,30y,50yr,80yr
River Rch & RM=RIVER-1,Reach-1         ,51.003
   25.18   27.74   29.24   31.13   32.87
River Rch & RM=RIVER-1,Reach-1         ,26
   37.23   41.04   43.27   46.08   48.66
Boundary for River Rch & Prof#=RIVER-1,Reach-1         , 1
Up Type= 0
Dn Type= 3
Dn Slope=.02
Boundary for River Rch & Prof#=RIVER-1,Reach-1         , 2
Up Type= 0
Dn Type= 3
Dn Slope=.02
Boundary for River Rch & Prof#=RIVER-1,Reach-1         , 3
Up Type= 0
Dn Type= 3
Dn Slope=.02
Boundary for River Rch & Prof#=RIVER-1,Reach-1         , 4
Up Type= 0
Dn Type= 3
Dn Slope=.02
Boundary for River Rch & Prof#=RIVER-1,Reach-1         , 5
Up Type= 0
Dn Type= 3
Dn Slope=.02
DSS Import GetInterval= 0
DSS Import GetPeak= 0
DSS Import FillOption= 0

--- bbc.g01 (geometry) ---

Geom Title=Imported Geom 01
Version=Version 3.0.1  Mar 2001

River Reach=RIVER-1         ,Reach-1
Reach XY= 2
              .5             .95              .5             .05

Type RM Length L Ch R = 1 ,51.003  ,3,3,3
#Sta/Elev= 6
     -10   71.63       0   71.63       3   69.03     8.5   69.03    11.7   71.63
    21.7   71.63
#Mann= 3 , 0 , 0
     -10    .035       0       0    .035       0    11.7    .035       0
#XS Ineff= 2 , 0
               0   71.63    11.7           71.63
Permanent Ineff=
       F       F
Bank Sta=0,11.7
XS Rating Curve= 0
Exp/Cntr=.3,.1

Type RM Length L Ch R = 1 ,51      ,50,50,50
#Sta/Elev= 14
   -20.8   78.24   -10.8   78.24    -7.8   76.04    -4.8   73.84    -1.8   71.64
       0   71.64     1.3   71.14     2.4   69.94     4.4   69.24     5.5   68.84
     6.5   68.84       7   69.94     9.2   71.64    19.2   71.64
#Mann= 3 , 0 , 0
   -20.8    .035       0       0    .035       0     9.2    .035       0
#XS Ineff= 2 , 0
               0   71.64     9.2           71.64
Permanent Ineff=
       F       F
Bank Sta=0,9.2
XS Rating Curve= 0
Exp/Cntr=.3,.1

Type RM Length L Ch R = 1 ,50      ,40,40,40
#Sta/Elev= 15
   -22.2   76.19   -12.2   76.19    -9.2   73.99    -6.2   71.79    -3.2   69.59
    -1.4   69.59     -.1   69.09       0   68.98       1   67.89       3   67.19
     4.1   66.79     5.1   66.79     5.6   67.89     7.8   68.99    17.8   68.99
#Mann= 3 , 0 , 0
   -22.2    .035       0    -1.4    .035       0     7.8    .035       0
Levee=-1,-1.4,69.59,-1,7.8,75,,
#XS Ineff= 2 , 0
            -1.4   69.59     7.8           68.99
Permanent Ineff=
       F       F
Bank Sta=-1.4,7.8
XS Rating Curve= 0
Exp/Cntr=.3,.1

Type RM Length L Ch R = 1 ,49.01   ,140,140,140
#Sta/Elev= 14
   -22.8   73.82   -12.8   73.82   -12.8   74.02   -12.6   74.02   -12.6   73.62
    -9.6   71.22    -9.6   68.92    -3.6   68.92     -.6   67.62       0    67.1
      .9   66.32     5.4   66.32     7.4   67.32    17.4   67.32
#Mann= 3 , 0 , 0
   -22.8    .035       0       0    .035       0     7.4    .035       0
Levee=-1,0,67.1,-1,7.4,70,,
#XS Ineff= 2 , 0
               0    67.1     7.4           67.32
Permanent Ineff=
       F       F
Bank Sta=0,7.4
XS Rating Curve= 0
Exp/Cntr=.3,.1

Type RM Length L Ch R = 1 ,46.02   ,20,20,20
#Sta/Elev= 6
     -10   66.97       0   66.97       0   65.67       8   65.67       8   66.77
      18   66.77
#Mann= 3 , 0 , 0
     -10    .035       0       0    .035       0       8    .035       0
Levee=-1,0,70,-1,8,70,,
#XS Ineff= 2 , 0
               0   66.97       8           66.77
Permanent Ineff=
       F       F
Bank Sta=0,8
XS Rating Curve= 0
Exp/Cntr=.3,.1

Type RM Length L Ch R = 1 ,46      ,16,16,16
#Sta/Elev= 9
     -10   63.27       0   63.27       0   61.77     2.7   61.77     2.7   63.27
     2.9   63.27     2.9   63.07     3.9   62.67    13.9   62.67
#Mann= 3 , 0 , 0
     -10    .035       0       0    .035       0     2.7    .035       0
Levee=-1,0,66,-1,2.7,66,,
#XS Ineff= 2 , 0
               0   63.27     2.7           63.27
Permanent Ineff=
       F       F
Bank Sta=0,2.7
XS Rating Curve= 0
Exp/Cntr=.3,.1

Type RM Length L Ch R = 1 ,45.034  ,4,4,4
#Sta/Elev= 11
   -11.5   60.72    -1.5   60.72       0   60.32       0   58.22     2.7   58.22
     2.7   60.42       3   60.42       3   60.12     3.5   60.12     5.8   58.32
    15.8   58.32
#Mann= 3 , 0 , 0
   -11.5    .035       0    -1.5    .035       0     2.7    .035       0
#XS Ineff= 2 , 0
       0    -1.5   60.72     2.7       0   58.22
Permanent Ineff=
       F       F
Bank Sta=-1.5,2.7
XS Rating Curve= 0
Exp/Cntr=.3,.1

Type RM Length L Ch R = 1 ,45.03   ,9,9,9
#Sta/Elev= 10
     -10   60.09       0   60.09       0   57.89       5   57.89       5   60.09
     5.3   60.09     5.3   59.39     5.8   59.39     6.4   58.39    16.4   58.39
#Mann= 3 , 0 , 0
     -10    .035       0       0    .035       0       5    .035       0
#XS Ineff= 2 , 0
               0   60.09       5           60.09
Permanent Ineff=
       F       F
Bank Sta=0,5
XS Rating Curve= 0
Exp/Cntr=.3,.1

Type RM Length L Ch R = 1 ,45.021  ,1,1,1
#Sta/Elev= 12
   -12.6   61.61    -2.6   61.61       0   59.44      .4   59.11      .8   57.81
     6.5   57.81     6.7   59.61     8.1   59.91     9.1   59.91    10.6   59.41
    11.2   58.21    21.2   58.21
#Mann= 3 , 0 , 0
   -12.6    .035       0    -2.6    .035       0     8.1    .035       0
#XS Ineff= 2 , 0
       0    -2.6   61.61     8.1       0   59.91
Permanent Ineff=
       F       F
Bank Sta=-2.6,8.1
XS Rating Curve= 0
Exp/Cntr=.3,.1

Type RM Length L Ch R = 1 ,45.02   ,20,20,20
#Sta/Elev= 14
   -12.6   61.44    -2.6   61.44       0   59.27      .4   58.94      .8   57.64
      .8   57.04     6.5   57.04     6.5   57.64     6.7   59.44     8.1   59.74
     9.1   59.74    10.6   59.24    11.2   58.04    21.2   58.04
#Mann= 3 , 0 , 0
   -12.6    .035       0    -2.6    .035       0     6.7    .035       0
#XS Ineff= 2 , 0
       0    -2.6   61.44     6.7       0   59.44
Permanent Ineff=
       F       F
Bank Sta=-2.6,6.7
XS Rating Curve= 0
Exp/Cntr=.3,.1

Type RM Length L Ch R = 1 ,45      ,50,50,50
#Sta/Elev= 11
   -10.9   58.72     -.9   58.72     -.4   58.32       0   58.32      .4   56.32
     4.9   56.32     5.5   58.32       7   58.82     7.5   58.82     7.7   58.62
    17.7   58.62
#Mann= 3 , 0 , 0
   -10.9    .035       0     -.9    .035       0       7    .035       0
#XS Ineff= 2 , 0
       0     -.9   58.72       7       0   58.82
Permanent Ineff=
       F       F
Bank Sta=-.9,7
XS Rating Curve= 0
Exp/Cntr=.3,.1

Type RM Length L Ch R = 1 ,44      ,21,21,21
#Sta/Elev= 11
   -10.9      57     -.9      57     -.4    56.6       0    56.6      .4    54.6
     4.9    54.6     5.5    56.6       7    57.4     7.5    57.4     7.7    57.2
    17.7    57.2
#Mann= 3 , 0 , 0
   -10.9    .035       0     -.9    .035       0       7    .035       0
Levee=-1,-.9,65,-1,7,65,,
#XS Ineff= 2 , 0
       0     -.9      57       7       0    57.4
Permanent Ineff=
       F       F
Bank Sta=-.9,7
XS Rating Curve= 0
Exp/Cntr=.3,.1

Type RM Length L Ch R = 1 ,43.029  ,2,2,2
#Sta/Elev= 6
     -10   56.28       0   56.28      .3   54.58     5.7   54.58       6   56.48
      16   56.48
#Mann= 3 , 0 , 0
     -10    .035       0       0    .035       0       6    .035       0
Levee=-1,0,60,-1,6,60,,
#XS Ineff= 2 , 0
               0   56.28       6           56.48
Permanent Ineff=
       F       F
Bank Sta=0,6
XS Rating Curve= 0
Exp/Cntr=.3,.1

Type RM Length L Ch R = 1 ,43.027  ,1,1,1
#Sta/Elev= 6
     -10   56.33       0   56.33       1   54.83     4.2   54.83     4.6   56.43
    14.6   56.43
#Mann= 3 , 0 , 0
     -10    .035       0       0    .035       0     4.6    .035       0
Levee=-1,0,60,-1,4.6,60,,
#XS Ineff= 2 , 0
               0   56.33     4.6           56.43
Permanent Ineff=
       F       F
Bank Sta=0,4.6
XS Rating Curve= 0
Exp/Cntr=.3,.1

Type RM Length L Ch R = 1 ,43.026  ,26,26,26
#Sta/Elev= 10
     -10   56.23       0   56.23       1   54.73       1   54.23     4.2   54.23
     4.2   54.73     4.6   56.33     5.6   56.33     6.4   55.93    16.4   55.93
#Mann= 3 , 0 , 0
     -10    .035       0       0    .035       0     4.6    .035       0
Levee=-1,0,60,-1,4.6,60,,
#XS Ineff= 2 , 0
               0   56.23     4.6           56.33
Permanent Ineff=
       F       F
Bank Sta=0,4.6
XS Rating Curve= 0
Exp/Cntr=.3,.1

Type RM Length L Ch R = 1 ,43      ,50,50,50
#Sta/Elev= 12
     -12   59.22      -9   58.42      -6   57.62      -3   56.82       0   55.62
      .4   54.32     2.2   53.62     5.2   53.62     7.5   55.22     8.5   55.22
     9.3   54.82    19.3   54.82
#Mann= 3 , 0 , 0
     -12    .035       0       0    .035       0     7.5    .035       0
Levee=-1,0,55.62,-1,7.5,60,,
#XS Ineff= 2 , 0
               0   55.62     7.5           55.22
Permanent Ineff=
       F       F
Bank Sta=0,7.5
XS Rating Curve= 0
Exp/Cntr=.3,.1

Type RM Length L Ch R = 1 ,42      ,50,50,50
#Sta/Elev= 12
     -12   57.46      -9   56.66      -6   55.86      -3   55.06       0   53.86
      .4   52.56     2.2   51.86     5.2   51.86     7.5   53.16     8.5   53.16
     9.3   52.76    19.3   52.76
#Mann= 3 , 0 , 0
     -12    .035       0       0    .035       0     7.5    .035       0
Levee=-1,0,53.86,-1,7.5,60,,
#XS Ineff= 2 , 0
               0   53.86     7.5           53.16
Permanent Ineff=
       F       F
Bank Sta=0,7.5
XS Rating Curve= 0
Exp/Cntr=.3,.1

Type RM Length L Ch R = 1 ,41      ,50,50,50
#Sta/Elev= 14
   -15.4   54.95    -5.4   54.95    -5.2   55.15    -4.9   55.15    -2.9   53.85
       0    52.3      .1   52.25     1.1   51.95     1.6   50.45     4.6   50.45
     7.6   52.45     8.2   52.45     8.4   52.25    18.4   52.25
#Mann= 3 , 0 , 0
   -15.4    .035       0    -4.9    .035       0     7.6    .035       0
#XS Ineff= 2 , 0
       0    -4.9   55.15     7.6       0   52.45
Permanent Ineff=
       F       F
Bank Sta=-4.9,7.6
XS Rating Curve= 0
Exp/Cntr=.3,.1

Type RM Length L Ch R = 1 ,40      ,2,2,2
#Sta/Elev= 15
   -15.4   54.49    -5.4   54.49    -5.2   54.69    -4.9   54.69      -4   54.06
    -2.9   53.29       0   51.65      .1   51.59     1.1   51.09     1.6   49.69
     4.6   49.69     7.6   51.79     8.2   51.79     8.4   51.59    18.4   51.59
#Mann= 3 , 0 , 0
   -15.4    .035       0    -4.9    .035       0     7.6    .035       0
#XS Ineff= 2 , 0
       0    -4.9   54.69     7.6       0   51.79
Permanent Ineff=
       F       F
Bank Sta=-4.9,7.6
XS Rating Curve= 0
Exp/Cntr=.3,.1

Type RM Length L Ch R = 1 ,39.048  ,1,1,1
#Sta/Elev= 14
   -14.4   53.74    -4.4   53.74    -4.2   53.94    -3.8   53.94      -3   53.34
       0   51.84       3   51.04     3.3   49.84     8.3   49.84     8.8   50.84
    10.1   51.84    10.6   51.84    10.9   51.64    20.9   51.64
#Mann= 3 , 0 , 0
   -14.4    .035       0    -3.8    .035       0    10.1    .035       0
#XS Ineff= 2 , 0
       0    -3.8   53.94    10.1       0   51.84
Permanent Ineff=
       F       F
Bank Sta=-3.8,10.1
XS Rating Curve= 0
Exp/Cntr=.3,.1

Type RM Length L Ch R = 1 ,39.047  ,14,14,14
#Sta/Elev= 16
   -14.4   53.74    -4.4   53.74    -4.2   53.94    -3.8   53.94      -3   53.34
       0   51.84       3   51.04     3.3   49.84     3.3   48.84     8.3   48.84
     8.3   49.84     8.8   50.84    10.1   51.84    10.6   51.84    10.9   51.64
    20.9   51.64
#Mann= 3 , 0 , 0
   -14.4    .035       0    -3.8    .035       0    10.1    .035       0
#XS Ineff= 2 , 0
       0    -3.8   53.94    10.1       0   51.84
Permanent Ineff=
       F       F
Bank Sta=-3.8,10.1
XS Rating Curve= 0
Exp/Cntr=.3,.1

Type RM Length L Ch R = 1 ,39.033  ,33,33,33
#Sta/Elev= 6
     -10   51.88       0   51.88      .3   49.18     5.3   49.18     5.6   51.88
    15.6   51.88
#Mann= 3 , 0 , 0
     -10    .035       0       0    .035       0     5.6    .035       0
#XS Ineff= 2 , 0
               0   51.88     5.6           51.88
Permanent Ineff=
       F       F
Bank Sta=0,5.6
XS Rating Curve= 0
Exp/Cntr=.3,.1

Type RM Length L Ch R = 1 ,39      ,50,50,50
#Sta/Elev= 16
    -9.9   54.61    -6.9   53.41    -3.9   52.21    -2.7   51.73     -.9   51.01
       0   50.11      .1   50.01      .1    50.1     2.1   48.01     5.1    48.1
     7.1   48.51     7.4   49.01     8.9   50.11     9.7   50.11    11.7   48.51
    21.7   48.51
#Mann= 3 , 0 , 0
    -9.9    .035       0       0    .035       0     8.9    .035       0
#XS Ineff= 2 , 0
               0   50.11     8.9           50.11
Permanent Ineff=
       F       F
Bank Sta=0,8.9
XS Rating Curve= 0
Exp/Cntr=.3,.1

Type RM Length L Ch R = 1 ,38      ,50,50,50
#Sta/Elev= 15
   -12.3   55.22    -9.3   54.32    -6.3   53.42    -3.3   52.52    -2.3   51.52
     -.3   49.52       0   49.22     1.7   47.52     4.7   47.52     6.7   48.02
       7   48.52     8.2   49.22       9   49.22      11   47.62      21   47.62
#Mann= 3 , 0 , 0
   -12.3    .035       0       0    .035       0     8.2    .035       0
#XS Ineff= 2 , 0
               0   49.22     8.2           49.22
Permanent Ineff=
       F       F
Bank Sta=0,8.2
XS Rating Curve= 0
Exp/Cntr=.3,.1

Type RM Length L Ch R = 1 ,37      ,50,50,50
#Sta/Elev= 13
      -9   49.17      -6   48.77      -3   48.37       0   47.97      .7   47.37
     2.7   46.27     4.3   46.27     4.8   46.87     5.5   47.37     5.8   48.77
     8.1   48.77     8.4   48.47    18.4   48.47
#Mann= 3 , 0 , 0
      -9    .035       0       0    .035       0     5.8    .035       0
#XS Ineff= 2 , 0
               0   47.97     5.8           48.77
Permanent Ineff=
       F       F
Bank Sta=0,5.8
XS Rating Curve= 0
Exp/Cntr=.3,.1

Type RM Length L Ch R = 1 ,36      ,50,50,50
#Sta/Elev= 12
      -6   47.68      -3   47.28       0   46.88      .7   46.28     2.7   45.18
     4.3   45.18     4.8   45.68     5.5   45.88     5.8   46.98     8.3   46.98
     8.5   46.78    18.5   46.78
#Mann= 3 , 0 , 0
      -6    .035       0       0    .035       0     5.8    .035       0
Levee=-1,0,50,-1,5.8,50,,
#XS Ineff= 2 , 0
               0   46.88     5.8           46.98
Permanent Ineff=
       F       F
Bank Sta=0,5.8
XS Rating Curve= 0
Exp/Cntr=.3,.1

Type RM Length L Ch R = 1 ,35      ,14,14,14
#Sta/Elev= 11
     -10   46.46       0   46.46      .6   44.76       1   44.76       1   44.46
       4   44.46       5   45.06       9   45.06     9.6   46.46    12.1   46.96
    22.1   46.96
#Mann= 3 , 0 , 0
     -10    .035       0       0    .035       0    12.1    .035       0
#XS Ineff= 2 , 0
               0   46.46    12.1           46.96
Permanent Ineff=
       F       F
Bank Sta=0,12.1
XS Rating Curve= 0
Exp/Cntr=.3,.1

Type RM Length L Ch R = 1 ,34.036  ,36,36,36
#Sta/Elev= 11
     -10   46.47       0   46.47      .7   44.47     1.1   44.47     1.1   44.17
     4.1   44.17     5.1   44.77     9.1   44.77     9.7   46.17    12.2   46.67
    22.2   46.67
#Mann= 3 , 0 , 0
     -10    .035       0       0    .035       0    12.2    .035       0
#XS Ineff= 2 , 0
               0   46.47    12.2           46.67
Permanent Ineff=
       F       F
Bank Sta=0,12.2
XS Rating Curve= 0
Exp/Cntr=.3,.1

Type RM Length L Ch R = 1 ,34      ,50,50,50
#Sta/Elev= 11
   -12.7    44.4    -2.7    44.4    -1.2    45.6       0    45.6     2.3    43.1
     6.3    43.1     6.3    44.3     7.5      45      10      45    11.2    44.2
    21.2    44.2
#Mann= 3 , 0 , 0
   -12.7    .035       0       0    .035       0     7.5    .035       0
Levee=-1,0,50,-1,7.5,50,,
#XS Ineff= 2 , 0
               0    45.6     7.5              45
Permanent Ineff=
       F       F
Bank Sta=0,7.5
XS Rating Curve= 0
Exp/Cntr=.3,.1

Type RM Length L Ch R = 1 ,33      ,22,22,22
#Sta/Elev= 6
     -10   44.27       0   44.27      .3   41.97     2.5   41.97     2.8   44.17
    12.8   44.17
#Mann= 3 , 0 , 0
     -10    .035       0       0    .035       0     2.8    .035       0
Levee=-1,0,50,-1,2.8,50,,
#XS Ineff= 2 , 0
               0   44.27     2.8           44.17
Permanent Ineff=
       F       F
Bank Sta=0,2.8
XS Rating Curve= 0
Exp/Cntr=.3,.1

Type RM Length L Ch R = 1 ,32.028  ,1,1,1
#Sta/Elev= 10
   -11.7   43.15    -1.7   43.15    -1.2   43.45       0   43.45      .4   41.15
     5.2   41.45     5.6   43.35     7.6   43.35       8   43.05      18   43.05
#Mann= 3 , 0 , 0
   -11.7    .035       0       0    .035       0     5.6    .035       0
#XS Ineff= 2 , 0
               0   43.45     5.6           43.35
Permanent Ineff=
       F       F
Bank Sta=0,5.6
XS Rating Curve= 0
Exp/Cntr=.3,.1

Type RM Length L Ch R = 1 ,32.027  ,27,27,27
#Sta/Elev= 12
   -11.7   43.15    -1.7   43.15    -1.2   43.45       0   43.45      .4   41.45
      .4   40.95     5.2   40.95     5.2   41.45     5.6   43.35     7.6   43.35
       8   43.05      18   43.05
#Mann= 3 , 0 , 0
   -11.7    .035       0       0    .035       0     5.6    .035       0
#XS Ineff= 2 , 0
               0   43.45     5.6           43.35
Permanent Ineff=
       F       F
Bank Sta=0,5.6
XS Rating Curve= 0
Exp/Cntr=.3,.1

Type RM Length L Ch R = 1 ,32      ,36,36,36
#Sta/Elev= 12
   -10.2   42.58     -.2   42.58     -.2   42.48       0   42.48      .3   40.58
     2.1   40.58     3.6   41.48     5.1   41.48     5.4   42.88       7   42.88
     7.6   42.48    17.6   42.48
#Mann= 3 , 0 , 0
   -10.2    .035       0       0    .035       0     5.4    .035       0
Levee=-1,0,51,-1,5.4,51,,
#XS Ineff= 2 , 0
       0       0   42.48     5.4       0   42.88
Permanent Ineff=
       F       F
Bank Sta=0,5.4
XS Rating Curve= 0
Exp/Cntr=.3,.1

Type RM Length L Ch R = 1 ,31.014  ,14,14,14
#Sta/Elev= 7
     -10   43.34       0   43.34      .6   40.84     3.6   40.24       6   40.24
     6.6   43.34    16.6   43.34
#Mann= 3 , 0 , 0
     -10    .035       0       0    .035       0     6.6    .035       0
#XS Ineff= 2 , 0
               0   43.34     6.6           43.34
Permanent Ineff=
       F       F
Bank Sta=0,6.6
XS Rating Curve= 0
Exp/Cntr=.3,.1

Type RM Length L Ch R = 1 ,31      ,29,29,29
#Sta/Elev= 9
     -10   43.22       0   43.22      .7   40.52     1.9   40.02     4.9   40.02
     5.5   43.32     5.7   43.32     5.7   43.72    15.7   43.72
#Mann= 3 , 0 , 0
     -10    .035       0       0    .035       0     5.7    .035       0
#XS Ineff= 2 , 0
               0   43.22     5.7           43.72
Permanent Ineff=
       F       F
Bank Sta=0,5.7
XS Rating Curve= 0
Exp/Cntr=.3,.1

Type RM Length L Ch R = 1 ,30.021  ,21,21,21
#Sta/Elev= 9
     -10   42.92       0   42.92      .7   39.92     1.9   39.42     5.1   39.42
     5.8   42.82       6   42.82       6   46.82      16   46.82
#Mann= 3 , 0 , 0
     -10    .035       0       0    .035       0       6    .035       0
#XS Ineff= 2 , 0
               0   42.92       6           46.82
Permanent Ineff=
       F       F
Bank Sta=0,6
XS Rating Curve= 0
Exp/Cntr=.3,.1

Type RM Length L Ch R = 1 ,30      ,18,18,18
#Sta/Elev= 10
     -10   41.54       0   41.54      .4   39.74     1.6   39.74     2.3   39.24
     4.7    39.2     5.2   42.54     5.4   42.54     5.4   42.94    15.4   42.94
#Mann= 3 , 0 , 0
     -10    .035       0       0    .035       0     5.4    .035       0
#XS Ineff= 2 , 0
               0   41.54     5.4           42.94
Permanent Ineff=
       F       F
Bank Sta=0,5.4
XS Rating Curve= 0
Exp/Cntr=.3,.1

Type RM Length L Ch R = 1 ,29.032  ,25,25,25
#Sta/Elev= 7
     -10   40.89       0   40.89      .4   39.39     3.9   39.39     5.4   38.99
     5.8   41.09    15.8   41.09
#Mann= 3 , 0 , 0
     -10    .035       0       0    .035       0     5.8    .035       0
Levee=-1,0,51,-1,5.8,51,,
#XS Ineff= 2 , 0
               0   40.89     5.8           41.09
Permanent Ineff=
       F       F
Bank Sta=0,5.8
XS Rating Curve= 0
Exp/Cntr=.3,.1

Type RM Length L Ch R = 1 ,29.007  ,1,1,1
#Sta/Elev= 10
   -10.2   40.02     -.2   40.02     -.2   40.22       0   40.22       0   39.02
     8.5   39.02     8.9   40.22     9.4   40.22    12.4   39.92    22.4   39.92
#Mann= 3 , 0 , 0
   -10.2    .035       0       0    .035       0     8.9    .035       0
Levee=-1,0,55,-1,8.9,55,,
#XS Ineff= 2 , 0
               0   40.22     8.9           40.22
Permanent Ineff=
       F       F
Bank Sta=0,8.9
XS Rating Curve= 0
Exp/Cntr=.3,.1

Type RM Length L Ch R = 1 ,29.006  ,5,5,5
#Sta/Elev= 11
   -10.2   40.02     -.2   40.02       0   40.22       0   39.02       0   38.02
     8.5   38.02     8.5   39.02     8.9   40.22     9.4   40.22    12.4   39.92
    22.4   39.92
#Mann= 3 , 0 , 0
   -10.2    .035       0       0    .035       0     8.9    .035       0
#XS Ineff= 2 , 0
               0   40.22     8.9           40.22
Permanent Ineff=
       F       F
Bank Sta=0,8.9
XS Rating Curve= 0
Exp/Cntr=.3,.1

Type RM Length L Ch R = 1 ,29.001  ,1,1,1
#Sta/Elev= 10
   -10.2   39.85     -.2   39.85     -.2   40.05       0   40.05       0   37.65
     8.5   37.65     8.9   40.05     9.4   40.05    12.4   39.75    22.4   39.75
#Mann= 3 , 0 , 0
   -10.2    .035       0       0    .035       0    12.4    .035       0
#XS Ineff= 2 , 0
               0   40.05    12.4           39.75
Permanent Ineff=
       F       F
Bank Sta=0,12.4
XS Rating Curve= 0
Exp/Cntr=.3,.1

Type RM Length L Ch R = 1 ,29      ,50,50,50
#Sta/Elev= 10
     -10   40.05       0   40.05       0   37.65       0   37.15     8.5   37.15
     8.5   37.65     8.9   40.05     9.4   40.05    12.4   39.75    22.4   39.75
#Mann= 3 , 0 , 0
     -10    .035       0       0    .035       0     8.9    .035       0
#XS Ineff= 2 , 0
               0   40.05     8.9           40.05
Permanent Ineff=
       F       F
Bank Sta=0,8.9
XS Rating Curve= 0
Exp/Cntr=.3,.1

Type RM Length L Ch R = 1 ,28      ,6,6,6
#Sta/Elev= 11
   -10.3   38.31     -.3   38.31     -.2   38.81       0   38.81       0   36.41
     1.3   36.41     1.7   36.01     2.9   36.01     5.3   36.81     5.7   39.01
    15.7   39.01
#Mann= 3 , 0 , 0
   -10.3    .035       0       0    .035       0     5.7    .035       0
#XS Ineff= 2 , 0
               0   38.81     5.7           39.01
Permanent Ineff=
       F       F
Bank Sta=0,5.7
XS Rating Curve= 0
Exp/Cntr=.3,.1

Type RM Length L Ch R = 1 ,27.044  ,44,44,44
#Sta/Elev= 9
     -10    38.4       0    38.4      .7    35.9      .9    35.9      .9    35.4
     3.9    35.4     6.9    36.6     7.5    38.5    17.5    38.5
#Mann= 3 , 0 , 0
     -10    .035       0       0    .035       0     7.5    .035       0
#XS Ineff= 2 , 0
               0    38.4     7.5            38.5
Permanent Ineff=
       F       F
Bank Sta=0,7.5
XS Rating Curve= 0
Exp/Cntr=.3,.1

Type RM Length L Ch R = 1 ,27      ,50,50,50
#Sta/Elev= 9
     -10    37.9       0    37.9      .7    35.4      .9    35.4      .9    34.7
     3.9    34.7     6.9    35.9     7.5    37.8    17.5    37.8
#Mann= 3 , 0 , 0
     -10    .035       0       0    .035       0     7.5    .035       0
#XS Ineff= 2 , 0
               0    37.9     7.5            37.8
Permanent Ineff=
       F       F
Bank Sta=0,7.5
XS Rating Curve= 0
Exp/Cntr=.3,.1

Type RM Length L Ch R = 1 ,26      ,50,50,50
#Sta/Elev= 12
     -10   37.16       0   37.16     1.6   36.26     2.1   34.36     5.3   34.36
     7.3   35.16     7.6   35.16     8.1   36.66       9   37.16     9.7   37.16
    10.7   36.36    20.7   36.36
#Mann= 3 , 0 , 0
     -10    .035       0       0    .035       0       9    .035       0
#XS Ineff= 2 , 0
               0   37.16       9           37.16
Permanent Ineff=
       F       F
Bank Sta=0,9
XS Rating Curve= 0
Exp/Cntr=.3,.1

Type RM Length L Ch R = 1 ,25      ,22,22,22
#Sta/Elev= 12
     -10   36.44       0   36.44     1.6   35.64     2.1   33.84     5.3   33.84
     7.3   34.64     7.6   34.64     8.1   36.14       9   36.64     9.7   36.64
    10.7   35.84    20.7   35.84
#Mann= 3 , 0 , 0
     -10    .035       0       0    .035       0       9    .035       0
#XS Ineff= 2 , 0
               0   36.44       9           36.64
Permanent Ineff=
       F       F
Bank Sta=0,9
XS Rating Curve= 0
Exp/Cntr=.3,.1

Type RM Length L Ch R = 1 ,24.028  ,28,28,28
#Sta/Elev= 6
     -10   36.39       0   36.39       0   33.39     9.8   33.39     9.8   36.39
    19.8   36.39
#Mann= 3 , 0 , 0
     -10    .035       0       0    .035       0     9.8    .035       0
#XS Ineff= 2 , 0
               0   36.39     9.8           36.39
Permanent Ineff=
       F       F
Bank Sta=0,9.8
XS Rating Curve= 0
Exp/Cntr=.3,.1

Type RM Length L Ch R = 1 ,24      ,10,10,10
#Sta/Elev= 6
     -10    36.2       0    36.2       0    33.4     9.4    33.4     9.4    36.2
    19.4    36.2
#Mann= 3 , 0 , 0
     -10    .035       0       0    .035       0     9.4    .035       0
#XS Ineff= 2 , 0
               0    36.2     9.4            36.2
Permanent Ineff=
       F       F
Bank Sta=0,9.4
XS Rating Curve= 0
Exp/Cntr=.3,.1

Type RM Length L Ch R = 1 ,23.04   ,11,11,11
#Sta/Elev= 6
     -10    36.2       0    36.2       0    33.3     9.8    33.3     9.8    36.2
    19.8    36.2
#Mann= 3 , 0 , 0
     -10    .035       0       0    .035       0     9.8    .035       0
#XS Ineff= 2 , 0
               0    36.2     9.8            36.2
Permanent Ineff=
       F       F
Bank Sta=0,9.8
XS Rating Curve= 0
Exp/Cntr=.3,.1

Type RM Length L Ch R = 1 ,23.029  ,29,29,29
#Sta/Elev= 12
     -10   35.15       0   35.15       1   34.45       1   32.95      11   32.95
    12.3   34.25    21.1   34.25    23.3   35.95    24.2   36.75    26.2   37.05
    26.7   37.45    36.7   37.45
#Mann= 3 , 0 , 0
     -10    .035       0       0    .035       0    12.3    .035       0
Levee=-1,0,41,-1,12.3,41,,
#XS Ineff= 2 , 0
               0   35.15    12.3           34.25
Permanent Ineff=
       F       F
Bank Sta=0,12.3
XS Rating Curve= 0
Exp/Cntr=.3,.1

Type RM Length L Ch R = 1 ,23      ,50,50,50
#Sta/Elev= 9
   -10.9   33.35     -.9   33.35     -.5   33.75       0   33.75      .3   32.55
    10.3   32.55    10.6   33.75    11.6   34.25    21.6   34.25
#Mann= 3 , 0 , 0
   -10.9    .035       0       0    .035       0    11.6    .035       0
Levee=-1,0,40,-1,11.6,40,,
#XS Ineff= 2 , 0
               0   33.75    11.6           34.25
Permanent Ineff=
       F       F
Bank Sta=0,11.6
XS Rating Curve= 0
Exp/Cntr=.3,.1

Type RM Length L Ch R = 1 ,22      ,50,50,50
#Sta/Elev= 9
   -10.8   33.26     -.8   33.26     -.5   33.56       0   33.56      .4   31.76
    12.4   31.76    12.8   33.56    13.8   34.26    23.8   34.26
#Mann= 3 , 0 , 0
   -10.8    .035       0       0    .035       0    13.8    .035       0
#XS Ineff= 2 , 0
               0   33.56    13.8           34.26
Permanent Ineff=
       F       F
Bank Sta=0,13.8
XS Rating Curve= 0
Exp/Cntr=.3,.1

Type RM Length L Ch R = 1 ,21      ,50,50,50
#Sta/Elev= 10
   -10.8   32.42     -.8   32.42     -.5   32.72       0   32.72      .4   30.92
    12.4   30.92    12.8   32.72    13.8   33.52    14.6   33.82    24.6   33.82
#Mann= 3 , 0 , 0
   -10.8    .035       0       0    .035       0    14.6    .035       0
#XS Ineff= 2 , 0
               0   32.72    14.6           33.82
Permanent Ineff=
       F       F
Bank Sta=0,14.6
XS Rating Curve= 0
Exp/Cntr=.3,.1

Type RM Length L Ch R = 1 ,20      ,50,50,50
#Sta/Elev= 13
   -11.1   31.97    -1.1   31.97     -.5   32.37       0   32.37      .5   30.77
     2.5   30.77     3.2   30.07     8.2   30.07     8.9   30.87    10.4   30.87
    10.8   32.77    11.8   32.27    21.8   32.27
#Mann= 3 , 0 , 0
   -11.1    .035       0       0    .035       0    10.8    .035       0
#XS Ineff= 2 , 0
       0       0   32.37    10.8       0   32.77
Permanent Ineff=
       F       F
Bank Sta=0,10.8
XS Rating Curve= 0
Exp/Cntr=.3,.1

Type RM Length L Ch R = 1 ,19      ,50,50,50
#Sta/Elev= 17
   -15.2   31.01    -5.2   31.01    -4.9   31.31      -2   31.31    -1.5   31.81
      -1   31.81     -.5   30.81       0   30.81      .5   28.81     2.5   28.81
       3   28.41       8   28.41     8.7   29.01    10.2   29.01    10.7   32.01
    11.5   32.41    21.5   32.41
#Mann= 3 , 0 , 0
   -15.2    .035       0      -1    .035       0    11.5    .035       0
Levee=-1,-1,41,-1,11.5,41,,
#XS Ineff= 2 , 0
              -1   31.81    11.5           32.41
Permanent Ineff=
       F       F
Bank Sta=-1,11.5
XS Rating Curve= 0
Exp/Cntr=.3,.1

Type RM Length L Ch R = 1 ,18      ,37,37,37
#Sta/Elev= 17
   -15.5   30.46    -5.5   30.46    -5.1   30.76    -2.1   30.76    -1.6   31.26
      -1   31.26     -.5   30.86       0   30.86      .5   29.46     2.5   29.46
       3   28.86       8   28.86     8.5   29.46      10   29.46    10.4   31.26
      11   31.46      21   31.46
#Mann= 3 , 0 , 0
   -15.5    .035       0      -1    .035       0      11    .035       0
Levee=-1,-1,40,-1,11,40,,
#XS Ineff= 2 , 0
              -1   31.26      11           31.46
Permanent Ineff=
       F       F
Bank Sta=-1,11
XS Rating Curve= 0
Exp/Cntr=.3,.1

Type RM Length L Ch R = 1 ,17.013  ,13,13,13
#Sta/Elev= 25
   -17.3   29.53    -7.3   29.53    -5.8   30.03    -1.8   30.03      -1   30.53
       0   30.53      .4   29.53      .8   29.53      .8   29.03     1.3   29.03
     1.3   29.53     1.5   29.53     1.5   29.23     2.8   29.23     2.8   28.73
     3.3   28.73     3.3   29.23     4.9   29.23     4.9   28.73     5.4   28.73
     5.4   29.23     6.6   29.23     7.1   30.53     7.3   30.63    17.3   30.63
#Mann= 3 , 0 , 0
   -17.3    .035       0       0    .035       0     7.3    .035       0
Levee=-1,0,40,-1,7.3,40,,
#XS Ineff= 2 , 0
               0   30.53     7.3           30.63
Permanent Ineff=
       F       F
Bank Sta=0,7.3
XS Rating Curve= 0
Exp/Cntr=.3,.1

Type RM Length L Ch R = 1 ,17      ,50,50,50
#Sta/Elev= 13
   -13.3   30.57    -3.3   30.57    -1.9   31.67       0   31.67     1.3   30.37
     2.9   29.27     4.5   28.57     6.6   28.57     8.6   29.27    10.7   30.47
      13   30.47    15.8   28.47    25.8   28.47
#Mann= 3 , 0 , 0
   -13.3    .035       0       0    .035       0    10.7    .035       0
Levee=-1,0,40,-1,10.7,40,,
#XS Ineff= 2 , 0
               0   31.67    10.7           30.47
Permanent Ineff=
       F       F
Bank Sta=0,10.7
XS Rating Curve= 0
Exp/Cntr=.3,.1

Type RM Length L Ch R = 1 ,16      ,50,50,50
#Sta/Elev= 13
   -13.3   30.08    -3.3   30.08    -1.9   31.18       0   31.18     1.3   29.88
     2.9   28.78     4.5   28.08     6.6   28.08     8.6   28.58    10.7   29.78
    13.1   29.78    16.2   27.38    26.2   27.38
#Mann= 3 , 0 , 0
   -13.3    .035       0       0    .035       0    10.7    .035       0
Levee=-1,0,40,-1,10.7,40,,
#XS Ineff= 2 , 0
               0   31.18    10.7           29.78
Permanent Ineff=
       F       F
Bank Sta=0,10.7
XS Rating Curve= 0
Exp/Cntr=.3,.1

Type RM Length L Ch R = 1 ,15      ,50,50,50
#Sta/Elev= 13
   -12.2   28.54    -2.2   28.54     -.9   29.74       0   29.74     2.5   28.34
     5.1   28.34     6.3   27.74     7.1   27.74     8.6   28.24    10.9   29.34
    13.4   29.34    15.6   27.94    25.6   27.94
#Mann= 3 , 0 , 0
   -12.2    .035       0       0    .035       0    10.9    .035       0
Levee=-1,0,40,-1,10.9,40,,
#XS Ineff= 2 , 0
               0   29.74    10.9           29.34
Permanent Ineff=
       F       F
Bank Sta=0,10.9
XS Rating Curve= 0
Exp/Cntr=.3,.1

Type RM Length L Ch R = 1 ,14      ,50,50,50
#Sta/Elev= 13
   -12.2   28.01    -2.2   28.01     -.9   29.21       0   29.21     2.5   27.81
     5.1   27.81     6.3   27.21     7.1   27.21     8.6   27.71    10.9   28.81
    13.4   28.81    15.6   27.41    25.6   27.41
#Mann= 3 , 0 , 0
   -12.2    .035       0       0    .035       0    10.9    .035       0
Levee=-1,0,40,-1,10.9,40,,
#XS Ineff= 2 , 0
               0   29.21    10.9           28.81
Permanent Ineff=
       F       F
Bank Sta=0,10.9
XS Rating Curve= 0
Exp/Cntr=.3,.1

Type RM Length L Ch R = 1 ,13      ,20,20,20
#Sta/Elev= 10
   -12.9   26.72    -2.9   26.72    -1.2   28.22       0   28.22     2.8   26.62
     6.8   26.62     9.6   28.12    12.1   28.12    14.1   26.52    24.2   26.51
#Mann= 3 , 0 , 0
   -12.9    .035       0       0    .035       0     9.6    .035       0
Levee=-1,0,40,-1,9.6,40,,
#XS Ineff= 2 , 0
               0   28.22     9.6           28.12
Permanent Ineff=
       F       F
Bank Sta=0,9.6
XS Rating Curve= 0
Exp/Cntr=.3,.1

Type RM Length L Ch R = 1 ,12.03   ,1,1,1
#Sta/Elev= 10
   -12.9   26.55    -2.9   26.55    -1.2   28.05       0   28.05     2.8   26.45
     6.8   26.45     9.6   27.95    12.4   27.95    14.6   26.05    24.6   26.05
#Mann= 3 , 0 , 0
   -12.9    .035       0       0    .035       0     9.6    .035       0
Levee=-1,0,40,-1,9.6,40,,
#XS Ineff= 2 , 0
               0   28.05     9.6           27.95
Permanent Ineff=
       F       F
Bank Sta=0,9.6
XS Rating Curve= 0
Exp/Cntr=.3,.1

Type RM Length L Ch R = 1 ,12.029  ,29,29,29
#Sta/Elev= 12
   -12.9   26.55    -2.9   26.55    -1.2   28.05       0   28.05     2.8   26.45
     2.8   25.45     6.8   25.45     6.8   26.45     9.6   27.95    12.4   27.95
    14.6   26.05    24.6   26.05
#Mann= 3 , 0 , 0
   -12.9    .035       0       0    .035       0     9.6    .035       0
Levee=-1,0,40,-1,9.6,40,,
#XS Ineff= 2 , 0
               0   28.05     9.6           27.95
Permanent Ineff=
       F       F
Bank Sta=0,9.6
XS Rating Curve= 0
Exp/Cntr=.3,.1

Type RM Length L Ch R = 1 ,12      ,50,50,50
#Sta/Elev= 12
     -13   26.34      -3   26.34    -1.2   27.64       0   27.64     2.4   26.04
     4.9   25.34     5.8   25.34     7.3   25.84    10.3   27.34    12.6   27.34
    15.1   25.74    25.1   25.74
#Mann= 3 , 0 , 0
     -13    .035       0       0    .035       0    10.3    .035       0
Levee=-1,0,40,-1,10.3,40,,
#XS Ineff= 2 , 0
               0   27.64    10.3           27.34
Permanent Ineff=
       F       F
Bank Sta=0,10.3
XS Rating Curve= 0
Exp/Cntr=.3,.1

Type RM Length L Ch R = 1 ,11      ,2,2,2
#Sta/Elev= 10
   -12.5   25.39    -2.5   25.39    -1.1   26.49       0   26.49       3   24.99
       7   24.99      10   26.49    12.4   26.49    14.6   24.69    24.6   24.69
#Mann= 3 , 0 , 0
   -12.5    .035       0       0    .035       0      10    .035       0
Levee=-1,0,40,-1,10,40,,
#XS Ineff= 2 , 0
               0   26.49      10           26.49
Permanent Ineff=
       F       F
Bank Sta=0,10
XS Rating Curve= 0
Exp/Cntr=.3,.1

Type RM Length L Ch R = 1 ,10.48   ,1,1,1
#Sta/Elev= 10
   -12.5   25.31    -2.5   25.31    -1.1   26.41       0   26.41       3   24.91
       7   24.91      10   26.41    12.4   26.41    14.6   24.61    24.6   24.61
#Mann= 3 , 0 , 0
   -12.5    .035       0       0    .035       0      10    .035       0
Levee=-1,0,40,-1,10,40,,
#XS Ineff= 2 , 0
               0   26.41      10           26.41
Permanent Ineff=
       F       F
Bank Sta=0,10
XS Rating Curve= 0
Exp/Cntr=.3,.1

Type RM Length L Ch R = 1 ,10.047  ,47,47,47
#Sta/Elev= 12
   -12.5   25.31    -2.5   25.31    -1.1   26.41       0   26.41       3   24.91
       3   23.91       7   23.91       7   24.91      10   26.41    12.4   26.41
    14.6   24.61    24.6   24.61
#Mann= 3 , 0 , 0
   -12.5    .035       0       0    .035       0      10    .035       0
Levee=-1,0,40,-1,10,40,,
#XS Ineff= 2 , 0
               0   26.41      10           26.41
Permanent Ineff=
       F       F
Bank Sta=0,10
XS Rating Curve= 0
Exp/Cntr=.3,.1

Type RM Length L Ch R = 1 ,10      ,50,50,50
#Sta/Elev= 12
   -12.4   24.38    -2.4   24.38     -.9   25.58       0   25.58     2.6   24.28
     2.8   23.68       6   23.68     6.3   24.18     9.3   25.68    11.7   25.68
    14.7   23.98    24.7   23.98
#Mann= 3 , 0 , 0
   -12.4    .035       0       0    .035       0     9.3    .035       0
Levee=-1,0,40,-1,9.3,40,,
#XS Ineff= 2 , 0
               0   25.58     9.3           25.68
Permanent Ineff=
       F       F
Bank Sta=0,9.3
XS Rating Curve= 0
Exp/Cntr=.3,.1

Type RM Length L Ch R = 1 ,9       ,32,32,32
#Sta/Elev= 10
   -12.3   23.79    -2.3   23.79      -1   24.99       0   24.99     2.5   23.19
     6.5   23.19     9.2   24.99    11.8   24.99    13.8   23.39    23.8   23.39
#Mann= 3 , 0 , 0
   -12.3    .035       0       0    .035       0     9.2    .035       0
Levee=-1,0,30,-1,9.2,30,,
#XS Ineff= 2 , 0
               0   24.99     9.2           24.99
Permanent Ineff=
       F       F
Bank Sta=0,9.2
XS Rating Curve= 0
Exp/Cntr=.3,.1

Type RM Length L Ch R = 1 ,8.018   ,1,1,1
#Sta/Elev= 10
   -12.3   23.53    -2.3   23.53      -1   24.73       0   24.73     2.5   23.13
     6.5   23.13     9.2   24.73    11.8   24.73    13.8   23.13    23.8   23.13
#Mann= 3 , 0 , 0
   -12.3    .035       0       0    .035       0     9.2    .035       0
Levee=-1,0,30,-1,9.2,30,,
#XS Ineff= 2 , 0
               0   24.73     9.2           24.73
Permanent Ineff=
       F       F
Bank Sta=0,9.2
XS Rating Curve= 0
Exp/Cntr=.3,.1

Type RM Length L Ch R = 1 ,8.017   ,17,17,17
#Sta/Elev= 12
   -12.3   23.53    -2.3   23.53      -1   24.73       0   24.73     2.5   23.13
     2.5   22.13     6.5   22.13     6.5   23.13     9.2   24.73    11.8   24.73
    13.8   23.13    23.8   23.13
#Mann= 3 , 0 , 0
   -12.3    .035       0       0    .035       0     9.2    .035       0
#XS Ineff= 2 , 0
               0   24.73     9.2           24.73
Permanent Ineff=
       F       F
Bank Sta=0,9.2
XS Rating Curve= 0
Exp/Cntr=.3,.1

Type RM Length L Ch R = 1 ,8       ,50,50,50
#Sta/Elev= 15
   -11.7    23.5    -1.7    23.5      -1    24.1       0    24.1       3    22.4
     4.7    22.4       6      22       7      22     7.8    22.6     8.7    22.6
    10.7    23.6    11.8    24.2    14.3    24.2    16.5    22.6    26.5    22.6
#Mann= 3 , 0 , 0
   -11.7    .035       0       0    .035       0    11.8    .035       0
Levee=-1,0,32,-1,11.8,32,,
#XS Ineff= 2 , 0
               0    24.1    11.8            24.2
Permanent Ineff=
       F       F
Bank Sta=0,11.8
XS Rating Curve= 0
Exp/Cntr=.3,.1

Type RM Length L Ch R = 1 ,7       ,36,36,36
#Sta/Elev= 9
     -10   23.61       0   23.61      .7   22.11     2.1   22.11     3.6   21.31
     6.6   21.31     9.6   21.93    10.2   23.31    20.2   23.31
#Mann= 3 , 0 , 0
     -10    .035       0       0    .035       0    10.2    .035       0
Levee=-1,0,30,-1,10.2,30,,
#XS Ineff= 2 , 0
               0   23.61    10.2           23.31
Permanent Ineff=
       F       F
Bank Sta=0,10.2
XS Rating Curve= 0
Exp/Cntr=.3,.1

Type RM Length L Ch R = 1 ,6.014   ,14,14,14
#Sta/Elev= 9
     -10   23.43       0   23.43      .7   21.93     2.1   21.93     3.6   21.13
     6.6   21.13     9.6   21.73    10.2   23.13    20.2   23.13
#Mann= 3 , 0 , 0
     -10    .035       0       0    .035       0    10.2    .035       0
Levee=-1,0,30,-1,10.2,30,,
#XS Ineff= 2 , 0
               0   23.43    10.2           23.13
Permanent Ineff=
       F       F
Bank Sta=0,10.2
XS Rating Curve= 0
Exp/Cntr=.3,.1

Type RM Length L Ch R = 1 ,6       ,17,17,17
#Sta/Elev= 8
     -10   24.67       0   24.67     1.7   20.97     2.9   21.27     6.1   21.27
     7.4   21.67     9.1   24.67    19.1   24.67
#Mann= 3 , 0 , 0
     -10    .035       0       0    .035       0     9.1    .035       0
#XS Ineff= 2 , 0
               0   24.67     9.1           24.67
Permanent Ineff=
       F       F
Bank Sta=0,9.1
XS Rating Curve= 0
Exp/Cntr=.3,.1

Type RM Length L Ch R = 1 ,5.033   ,1,1,1
#Sta/Elev= 10
   -12.8   21.37    -2.8   21.37    -1.5   22.47       0   22.47     3.2   20.67
     7.2   20.67    10.4   22.47    12.8   22.47    14.3   20.67    24.3   20.67
#Mann= 3 , 0 , 0
   -12.8    .035       0       0    .035       0    10.4    .035       0
Levee=-1,0,30,-1,10.4,30,,
#XS Ineff= 2 , 0
               0   22.47    10.4           22.47
Permanent Ineff=
       F       F
Bank Sta=0,10.4
XS Rating Curve= 0
Exp/Cntr=.3,.1

Type RM Length L Ch R = 1 ,5.032   ,32,32,32
#Sta/Elev= 12
   -12.8   21.37    -2.8   21.37    -1.5   22.47       0   22.47     3.2   20.67
     3.2   19.67     7.2   19.67     7.2   20.67    10.4   22.47    12.8   22.47
    14.3   20.67    24.3   20.67
#Mann= 3 , 0 , 0
   -12.8    .035       0       0    .035       0    10.4    .035       0
#XS Ineff= 2 , 0
               0   22.47    10.4           22.47
Permanent Ineff=
       F       F
Bank Sta=0,10.4
XS Rating Curve= 0
Exp/Cntr=.3,.1

Type RM Length L Ch R = 1 ,5       ,50,50,50
#Sta/Elev= 10
   -12.8   20.38    -2.8   20.38    -1.5   21.48       0   21.48     3.2   19.58
     7.2   19.58    10.4   21.48    12.7   21.48    14.5   19.88    24.5   19.88
#Mann= 3 , 0 , 0
   -12.8    .035       0       0    .035       0    10.4    .035       0
Levee=-1,0,32,-1,10.4,32,,
#XS Ineff= 2 , 0
               0   21.48    10.4           21.48
Permanent Ineff=
       F       F
Bank Sta=0,10.4
XS Rating Curve= 0
Exp/Cntr=.3,.1

Type RM Length L Ch R = 1 ,4       ,50,50,50
#Sta/Elev= 15
     -13   19.53      -3   19.53    -1.5   20.93    -1.1   21.33       0   21.33
       2   20.13       5   18.93     6.3   18.93     6.5   19.13     7.2   19.13
     7.4   19.43     9.9   20.73    12.1   20.73    13.1   19.73    23.1   19.73
#Mann= 3 , 0 , 0
     -13    .035       0       0    .035       0     9.9    .035       0
Levee=-1,0,23,-1,9.9,22,,
#XS Ineff= 2 , 0
               0   21.33     9.9           20.73
Permanent Ineff=
       F       F
Bank Sta=0,9.9
XS Rating Curve= 0
Exp/Cntr=.3,.1

Type RM Length L Ch R = 1 ,3       ,40,40,40
#Sta/Elev= 11
   -12.7   19.29    -2.7   19.29      -1   20.79       0   20.79      .6   20.29
     2.9   18.69     6.9   18.69     9.4   20.29    11.6   20.29    13.6   18.89
    23.6   18.89
#Mann= 3 , 0 , 0
   -12.7    .035       0       0    .035       0     9.4    .035       0
Levee=-1,0,22,-1,9.4,22,,
#XS Ineff= 2 , 0
               0   20.79     9.4           20.29
Permanent Ineff=
       F       F
Bank Sta=0,9.4
XS Rating Curve= 0
Exp/Cntr=.3,.1

Type RM Length L Ch R = 1 ,2.01    ,10,10,10
#Sta/Elev= 11
   -12.7   18.83    -2.7   18.83      -1   20.33       0   20.33      .6   19.73
     2.9   18.03     6.9   18.03     9.4   19.73    11.6   19.73    13.6   18.33
    23.6   18.33
#Mann= 3 , 0 , 0
   -12.7    .035       0       0    .035       0     9.4    .035       0
Levee=-1,0,20.33,-1,9.4,22,,
#XS Ineff= 2 , 0
               0   20.33     9.4           19.73
Permanent Ineff=
       F       F
Bank Sta=0,9.4
XS Rating Curve= 0
Exp/Cntr=.3,.1

Type RM Length L Ch R = 1 ,2       ,50,50,50
#Sta/Elev= 13
   -12.9   18.21    -2.9   18.21     -.9   19.81       0   19.81      .7   19.11
     2.9   17.51     5.1   17.51     6.4   17.11       7   17.11    10.5   19.71
    12.7   19.71    14.8   18.01    24.8   18.01
#Mann= 3 , 0 , 0
   -12.9    .035       0       0    .035       0    10.5    .035       0
Levee=-1,0,31,-1,10.5,31,,
#XS Ineff= 2 , 0
               0   19.81    10.5           19.71
Permanent Ineff=
       F       F
Bank Sta=0,10.5
XS Rating Curve= 0
Exp/Cntr=.3,.1

Type RM Length L Ch R = 1 ,1       ,50,50,50
#Sta/Elev= 13
   -13.1   17.69    -3.1   17.69     -.9   19.49       0   19.49      .7   18.79
     2.7   17.29     4.9   17.29     6.2   16.89     6.8   16.89    10.3   19.29
    12.5   19.29    14.6   17.59    24.6   17.59
#Mann= 3 , 0 , 0
   -13.1    .035       0       0    .035       0    10.3    .035       0
#XS Ineff= 2 , 0
               0   19.49    10.3           19.29
Permanent Ineff=
       F       F
Bank Sta=0,10.3
XS Rating Curve= 0
Exp/Cntr=.3,.1

Type RM Length L Ch R = 1 ,0       ,0,0,0
#Sta/Elev= 6
     -10   18.86       0   18.86       0   16.16     6.5   16.16     6.5   18.86
    16.5   18.86
#Mann= 3 , 0 , 0
     -10    .035       0       0    .035       0     6.5    .035       0
#XS Ineff= 2 , 0
               0   18.86     6.5           18.86
Permanent Ineff=
       F       F
Bank Sta=0,6.5
XS Rating Curve= 0
Exp/Cntr=.3,.1

Chan Stop Cuts=-1
