--- SIN.prj (project) ---

Proj Title=SIN
Current Plan=p01
Default Exp/Contr=.3,.1
SI Units
Geom File=g01
Flow File=f01
Plan File=p01
Y Axis Title=Elevation
X Axis Title(PF)=Main Channel Distance
X Axis Title(XS)=Station
BEGIN DESCRIPTION:
           BACK WATER COMPUTATION
      APPLICATION OF HEC-2 BY Samju Construction Engineering
      sinsan-ch: 10,20,30,50,80 yr
END DESCRIPTION:
DSS Export Rating Curves= 0
DSS Export Rating Curve Sorted= 0
DSS Export Volume Flow Curves= 0
DXF OffsetX= 0
DXF OffsetY= 0
DXF ScaleX= 1
DXF ScaleY= 10

--- SIN.p01 (plan) ---

Plan Title=Imported Plan 01
Version=Version 3.0.1  Mar 2001
Short Identifier=Imported Pla
Geom File=g01
Flow File=f01
Subcritical Flow
K Sum by GR= 0
Std Step Tol= 0.003
Critical Tol= 0.003
Num of Std Step Trials= 20
Max Error Tol= 0.1
Flow Tol Ratio= 0.001
Split Flow NTrial= 30
Split Flow Tol= 0.02
Split Flow Ratio= 0.02
Log Output Level= 0
Friction Slope Method= 1
Unsteady Friction Slope Method= 2
Parabolic Critical Depth
Global Vel Dist= 0 , 0 , 0
Global Log Level= 0
CheckData=True
Encroach Param=-1 ,0,0, 0
Computation Interval=1HOUR
Output Interval=1HOUR
Run HTab= 0
Run UNet= 0
Run PostProcess= 0
UNET Theta= 1
UNET ZTol= 0.02
UNET ZSATol= 0.1
UNET MxIter= 20
UNET MaxInSteps= 20
UNET DtIC= 0
UNET DtMin= 0
UNET MaxCRTS= 20
UNET WFStab= 2
UNET SFStab= 1
UNET WFX= 1
UNET SFX= 1
UNET Convert EG Bridges=-1
UNET Use Existing IB Tables=-1
Instantaneous Interval=1HOUR
Write IC File= 0
Write Velocity= 0
Write Detailed= 0

--- SIN.f01 (steady flow) ---

Flow Title=Imported Flow 01
Version=Version 3.0.1  Mar 2001
Number of Profiles= 5
Profile Names=10YR,20YR,30YR,50YR,80YR
River Rch & RM=RIVER-1,Reach-1         ,2589.00
     9.9    10.9   11.48   12.22    12.9
River Rch & RM=RIVER-1,Reach-1         ,2000.00
   21.98   24.22   25.52   27.17   28.69
River Rch & RM=RIVER-1,Reach-1         ,750.00
   28.19   31.07   32.75   34.88   36.83
Boundary for River Rch & Prof#=RIVER-1,Reach-1         , 1
Up Type= 0
Dn Type= 3
Dn Slope=.028
Boundary for River Rch & Prof#=RIVER-1,Reach-1         , 2
Up Type= 0
Dn Type= 3
Dn Slope=.028
Boundary for River Rch & Prof#=RIVER-1,Reach-1         , 3
Up Type= 0
Dn Type= 3
Dn Slope=.028
Boundary for River Rch & Prof#=RIVER-1,Reach-1         , 4
Up Type= 0
Dn Type= 3
Dn Slope=.028
Boundary for River Rch & Prof#=RIVER-1,Reach-1         , 5
Up Type= 0
Dn Type= 3
Dn Slope=.028
DSS Import GetInterval= 0
DSS Import GetPeak= 0
DSS Import FillOption= 0

--- SIN.g01 (geometry) ---

Geom Title=Imported Geom 01
Version=Version 3.0.1  Mar 2001

River Reach=RIVER-1         ,Reach-1
Reach XY= 2
              .5             .95              .5             .05

Type RM Length L Ch R = 1 ,2589.00 ,20,20,20
BEGIN DESCRIPTION:
51.02
END DESCRIPTION:
#Sta/Elev= 9
     -10  122.66       0  122.66      .8  120.96     3.3  120.96     5.1  122.06
     7.1  123.06     8.6  123.86    11.6  124.46    21.6  124.46
#Mann= 3 , 0 , 0
     -10    .035       0       0    .035       0    11.6    .035       0
#XS Ineff= 2 , 0
               0     130    11.6             130
Permanent Ineff=
       F       F
#Block Obstruct= 2 , 0
                            11.6
Bank Sta=0,11.6
XS Rating Curve= 0
Exp/Cntr=.3,.1

Type RM Length L Ch R = 1 ,2569.00 ,1,1,1
BEGIN DESCRIPTION:
51.019
END DESCRIPTION:
#Sta/Elev= 12
   -14.5  122.91    -4.5  122.91      -2  122.71       0  122.51     1.3  121.51
     1.5  121.51     2.8  121.01     4.1  121.01     5.7  121.71     7.3  122.31
       8  122.91      11  123.21
#Mann= 3 , 0 , 0
   -14.5    .035       0      -2    .035       0     7.3    .035       0
#XS Ineff= 2 , 0
              -2     130     7.3             130
Permanent Ineff=
       F       F
#Block Obstruct= 2 , 0
                             7.3
Bank Sta=-2,7.3
XS Rating Curve= 0
Exp/Cntr=.3,.1

Type RM Length L Ch R = 1 ,2568.00 ,18,18,18
BEGIN DESCRIPTION:
51.018
END DESCRIPTION:
#Sta/Elev= 14
   -14.5  122.91    -4.5  122.91      -2  122.71       0  122.51     1.3  121.51
     1.5  121.51     2.8  121.01     2.8  120.01     4.1  120.01     4.1  121.01
     5.7  121.72     7.3  122.31       8  122.91      11  123.21
#Mann= 3 , 0 , 0
   -14.5    .035       0      -2    .035       0     7.3    .035       0
#XS Ineff= 2 , 0
              -2     125     7.3             125
Permanent Ineff=
       F       F
#Block Obstruct= 2 , 0
                             7.3
Bank Sta=-2,7.3
XS Rating Curve= 0
Exp/Cntr=.3,.1

Type RM Length L Ch R = 1 ,2550.00 ,50,50,50
BEGIN DESCRIPTION:
51
END DESCRIPTION:
#Sta/Elev= 12
   -14.5  121.51    -4.5  121.51      -2  121.31       0  121.11     1.3  120.11
     1.5  120.11     2.8  121.11     4.1  121.11     5.7  122.11     7.3  122.91
       8  123.51      11  123.81
#Mann= 3 , 0 , 0
   -14.5    .035       0       0    .035       0     2.8    .035       0
#XS Ineff= 2 , 0
               0     125     2.8             125
Permanent Ineff=
       F       F
#Block Obstruct= 2 , 0
                             2.8
Bank Sta=0,2.8
XS Rating Curve= 0
Exp/Cntr=.3,.1

Type RM Length L Ch R = 1 ,2500.00 ,14,14,14
BEGIN DESCRIPTION:
50
END DESCRIPTION:
#Sta/Elev= 10
   -14.7  117.18    -4.7  117.18    -3.9  117.88       0  117.88     3.2  115.98
     5.1  115.98     7.8  117.98     9.2  117.98     9.8  117.38    19.8  117.38
#Mann= 3 , 0 , 0
   -14.7    .035       0       0    .035       0     7.8    .035       0
#XS Ineff= 2 , 0
               0     125     7.8             125
Permanent Ineff=
       F       F
#Block Obstruct= 2 , 0
                             7.8
Bank Sta=0,7.8
XS Rating Curve= 0
Exp/Cntr=.3,.1

Type RM Length L Ch R = 1 ,2486.00 ,26,26,26
BEGIN DESCRIPTION:
49.036
END DESCRIPTION:
#Sta/Elev= 8
   -18.3  116.88    -8.3  116.88      -6  118.58       0  118.58       0  116.88
       2  116.88       2  118.58      12  118.58
#Mann= 3 , 0 , 0
   -18.3    .035       0       0    .035       0       2    .035       0
#XS Ineff= 2 , 0
               0     125       2             125
Permanent Ineff=
       F       F
#Block Obstruct= 2 , 0
                               2
Bank Sta=0,2
XS Rating Curve= 0
Exp/Cntr=.3,.1

Type RM Length L Ch R = 1 ,2460.00 ,1,1,1
BEGIN DESCRIPTION:
49.01
END DESCRIPTION:
#Sta/Elev= 9
   -13.7  116.93    -3.7  116.93       0  116.93     1.1  116.03     1.3  116.03
     2.6  115.53     4.2  115.53     5.9  116.03    15.9  116.03
#Mann= 3 , 0 , 0
   -13.7    .035       0       0    .035       0     5.9    .035       0
#XS Ineff= 2 , 0
               0     125     5.9             125
Permanent Ineff=
       F       F
#Block Obstruct= 2 , 0
                             5.9
Bank Sta=0,5.9
XS Rating Curve= 0
Exp/Cntr=.3,.1

Type RM Length L Ch R = 1 ,2459.00 ,9,9,9
BEGIN DESCRIPTION:
49.009
END DESCRIPTION:
#Sta/Elev= 11
   -13.7  114.37    -3.7  114.37       0  116.93     1.1  116.03     1.3  116.03
     2.6  115.53     2.6  114.33     4.2  114.33     4.2  115.53     5.9  116.03
    15.9  116.03
#Mann= 3 , 0 , 0
   -13.7    .035       0       0    .035       0     5.9    .035       0
#XS Ineff= 2 , 0
               0     125     5.9             125
Permanent Ineff=
       F       F
#Block Obstruct= 2 , 0
                             5.9
Bank Sta=0,5.9
XS Rating Curve= 0
Exp/Cntr=.3,.1

Type RM Length L Ch R = 1 ,2450.00 ,21,21,21
BEGIN DESCRIPTION:
49
END DESCRIPTION:
#Sta/Elev= 9
   -13.7  116.26    -3.7  116.26       0  116.26     1.1  115.36     1.3  115.36
     2.6  114.36     4.2  114.36     5.9  115.36    15.9  115.36
#Mann= 3 , 0 , 0
   -13.7    .035       0       0    .035       0     5.9    .035       0
#XS Ineff= 2 , 0
               0     125     5.9             125
Permanent Ineff=
       F       F
#Block Obstruct= 2 , 0
                             5.9
Bank Sta=0,5.9
XS Rating Curve= 0
Exp/Cntr=.3,.1

Type RM Length L Ch R = 1 ,2429.00 ,1,1,1
BEGIN DESCRIPTION:
48.029
END DESCRIPTION:
#Sta/Elev= 9
   -13.7  114.99    -3.7  114.99       0  114.99     1.1  114.09     1.3  114.09
     2.6  113.69     4.2  113.69     5.9  114.09    15.9  114.09
#Mann= 3 , 0 , 0
   -13.7    .035       0       0    .035       0     5.9    .035       0
#XS Ineff= 2 , 0
               0     125     5.9             125
Permanent Ineff=
       F       F
#Block Obstruct= 2 , 0
                             5.9
Bank Sta=0,5.9
XS Rating Curve= 0
Exp/Cntr=.3,.1

Type RM Length L Ch R = 1 ,2428.00 ,28,28,28
BEGIN DESCRIPTION:
48.028
END DESCRIPTION:
#Sta/Elev= 11
   -13.7  114.99    -3.7  114.99       0  114.99     1.1  114.09     1.3  114.09
     2.6  113.69     2.6  112.49     4.2  112.49     4.2  113.69     5.9  114.09
    15.9  114.09
#Mann= 3 , 0 , 0
   -13.7    .035       0       0    .035       0     2.6    .035       0
#XS Ineff= 2 , 0
               0     125     2.6             125
Permanent Ineff=
       F       F
#Block Obstruct= 2 , 0
                             2.6
Bank Sta=0,2.6
XS Rating Curve= 0
Exp/Cntr=.3,.1

Type RM Length L Ch R = 1 ,2400.00 ,2,2,2
BEGIN DESCRIPTION:
48
END DESCRIPTION:
#Sta/Elev= 13
   -15.1  113.82    -5.1  113.82    -4.9  114.02    -4.7  114.02    -3.7  113.72
       0  113.72       0  112.12       2  112.12       2  113.72     2.3  113.72
     2.9  113.32     4.7  112.32    14.7  112.32
#Mann= 3 , 0 , 0
   -15.1    .035       0       0    .035       0       2    .035       0
#XS Ineff= 2 , 0
               0     125       2             125
Permanent Ineff=
       F       F
#Block Obstruct= 2 , 0
                               2
Bank Sta=0,2
XS Rating Curve= 0
Exp/Cntr=.3,.1

Type RM Length L Ch R = 1 ,2398.00 ,32,32,32
BEGIN DESCRIPTION:
47.048
END DESCRIPTION:
#Sta/Elev= 13
   -15.1  113.86    -5.1  113.86    -4.9  114.06    -4.7  114.06    -3.7  113.76
       0  113.76       0  112.16       2  112.16       2  113.76     2.3  113.76
     2.9  113.36     4.7  112.36    14.7  112.36
#Mann= 3 , 0 , 0
   -15.1    .035       0       0    .035       0       2    .035       0
#XS Ineff= 2 , 0
               0     125       2             125
Permanent Ineff=
       F       F
#Block Obstruct= 2 , 0
                               2
Bank Sta=0,2
XS Rating Curve= 0
Exp/Cntr=.3,.1

Type RM Length L Ch R = 1 ,2366.00 ,16,16,16
BEGIN DESCRIPTION:
47.016
END DESCRIPTION:
#Sta/Elev= 8
     -10  113.19       0  113.19       0  111.39     2.1  111.39     2.1  113.19
     7.1  113.19    12.6  107.69    22.6  107.69
#Mann= 3 , 0 , 0
     -10    .035       0       0    .035       0     2.1    .035       0
#XS Ineff= 2 , 0
               0     120     2.1             120
Permanent Ineff=
       F       F
#Block Obstruct= 2 , 0
                             2.1
Bank Sta=0,2.1
XS Rating Curve= 0
Exp/Cntr=.3,.1

Type RM Length L Ch R = 1 ,2350.00 ,24,24,24
BEGIN DESCRIPTION:
47
END DESCRIPTION:
#Sta/Elev= 13
   -15.6  113.75    -5.6  113.75    -5.3  114.05    -3.9  112.75    -3.9  112.35
    -3.5  112.35    -3.5  112.75    -2.5  113.35       0  113.35     2.8  111.55
       5  111.55     7.8  113.35    10.8  113.35
#Mann= 3 , 0 , 0
   -15.6    .035       0       0    .035       0     7.8    .035       0
#XS Ineff= 2 , 0
               0     120     7.8             120
Permanent Ineff=
       F       F
#Block Obstruct= 2 , 0
                             7.8
Bank Sta=0,7.8
XS Rating Curve= 0
Exp/Cntr=.3,.1

Type RM Length L Ch R = 1 ,2326.00 ,16,16,16
BEGIN DESCRIPTION:
46.026
END DESCRIPTION:
#Sta/Elev= 13
   -15.6  113.38    -5.6  113.38    -5.3  113.68    -3.9  112.38    -3.9  111.98
    -3.5  111.98    -3.5  112.38    -2.5  112.98       0  112.98     2.8  111.18
       5  111.18     7.8  112.98    10.8  112.98
#Mann= 3 , 0 , 0
   -15.6    .035       0       0    .035       0     7.8    .035       0
#XS Ineff= 2 , 0
               0     120     7.8             120
Permanent Ineff=
       F       F
#Block Obstruct= 2 , 0
                             7.8
Bank Sta=0,7.8
XS Rating Curve= 0
Exp/Cntr=.3,.1

Type RM Length L Ch R = 1 ,2310.00 ,1,1,1
BEGIN DESCRIPTION:
46.01
END DESCRIPTION:
#Sta/Elev= 8
     -10  112.85       0  112.85       0  112.65     1.5  112.15     1.5  110.65
     3.7  110.65     3.7  112.15    13.7  112.15
#Mann= 3 , 0 , 0
     -10    .035       0       0    .035       0     3.7    .035       0
#XS Ineff= 2 , 0
               0     120     3.7             120
Permanent Ineff=
       F       F
#Block Obstruct= 2 , 0
                             3.7
Bank Sta=0,3.7
XS Rating Curve= 0
Exp/Cntr=.3,.1

Type RM Length L Ch R = 1 ,2309.00 ,9,9,9
BEGIN DESCRIPTION:
46.009
END DESCRIPTION:
#Sta/Elev= 10
     -10  112.85       0  112.85       0  112.65     1.5  112.15     1.5  110.65
     1.5  109.85     3.7  109.85     3.7  110.65     3.7  112.15    13.7  112.15
#Mann= 3 , 0 , 0
     -10    .035       0       0    .035       0     3.7    .035       0
#XS Ineff= 2 , 0
               0     120     3.7             120
Permanent Ineff=
       F       F
#Block Obstruct= 2 , 0
                             3.7
Bank Sta=0,3.7
XS Rating Curve= 0
Exp/Cntr=.3,.1

Type RM Length L Ch R = 1 ,2300.00 ,50,50,50
BEGIN DESCRIPTION:
46
END DESCRIPTION:
#Sta/Elev= 12
   -14.6  110.15    -4.6  110.15      -3  111.55      -3  111.75       0  111.75
       0  111.55     2.7  108.55       4  108.55     5.9  110.35     6.3  110.35
     6.9  109.95    16.9  109.95
#Mann= 3 , 0 , 0
   -14.6    .035       0       0    .035       0     5.9    .035       0
#XS Ineff= 2 , 0
               0     120     5.9             120
Permanent Ineff=
       F       F
#Block Obstruct= 2 , 0
                             5.9
Bank Sta=0,5.9
XS Rating Curve= 0
Exp/Cntr=.3,.1

Type RM Length L Ch R = 1 ,2250.00 ,50,50,50
BEGIN DESCRIPTION:
45
END DESCRIPTION:
#Sta/Elev= 10
   -13.8  108.41    -3.8  108.41      -3  109.11       0  109.11     2.2  106.41
     3.7  106.41     5.4  108.61     5.7  108.61     5.9  108.41    15.9  108.41
#Mann= 3 , 0 , 0
   -13.8    .035       0       0    .035       0     5.4    .035       0
#XS Ineff= 2 , 0
               0     115     5.4             115
Permanent Ineff=
       F       F
#Block Obstruct= 2 , 0
                             5.4
Bank Sta=0,5.4
XS Rating Curve= 0
Exp/Cntr=.3,.1

Type RM Length L Ch R = 1 ,2200.00 ,33,33,33
BEGIN DESCRIPTION:
44
END DESCRIPTION:
#Sta/Elev= 10
   -13.8  106.71    -3.8  106.71      -3  107.41       0  107.41     2.2  105.51
     3.7  105.51     5.4  106.91     5.7  106.91     5.9  106.71    15.9  106.71
#Mann= 3 , 0 , 0
   -13.8    .035       0       0    .035       0     5.4    .035       0
#XS Ineff= 2 , 0
               0     115     5.4             115
Permanent Ineff=
       F       F
#Block Obstruct= 2 , 0
                             5.4
Bank Sta=0,5.4
XS Rating Curve= 0
Exp/Cntr=.3,.1

Type RM Length L Ch R = 1 ,2167.00 ,17,17,17
BEGIN DESCRIPTION:
43.017
END DESCRIPTION:
#Sta/Elev= 10
   -14.4  105.45    -4.4  105.45      -3  106.85       0  106.85     1.5  105.35
     3.7  105.35     5.8  106.85     6.1  106.85     6.3  106.65    16.3  106.65
#Mann= 3 , 0 , 0
   -14.4    .035       0       0    .035       0     5.8    .035       0
#XS Ineff= 2 , 0
               0     115     5.8             115
Permanent Ineff=
       F       F
#Block Obstruct= 2 , 0
                             5.8
Bank Sta=0,5.8
XS Rating Curve= 0
Exp/Cntr=.3,.1

Type RM Length L Ch R = 1 ,2150.00 ,50,50,50
BEGIN DESCRIPTION:
43
END DESCRIPTION:
#Sta/Elev= 10
   -14.4  104.95    -4.4  104.95      -3  106.35       0  106.35     1.5  105.05
     3.7  105.05     5.8  106.35     6.1  106.35     6.3  106.15    16.3  106.15
#Mann= 3 , 0 , 0
   -14.4    .035       0       0    .035       0     5.8    .035       0
#XS Ineff= 2 , 0
               0     110     5.8             110
Permanent Ineff=
       F       F
#Block Obstruct= 2 , 0
                             5.8
Bank Sta=0,5.8
XS Rating Curve= 0
Exp/Cntr=.3,.1

Type RM Length L Ch R = 1 ,2100.00 ,50,50,50
BEGIN DESCRIPTION:
42
END DESCRIPTION:
#Sta/Elev= 10
   -14.5  104.11    -4.5  104.11      -3  105.51       0  105.51     1.6  104.41
     3.2  104.41     5.8  106.11     6.2  106.11     6.4  105.91    16.4  105.91
#Mann= 3 , 0 , 0
   -14.5    .035       0       0    .035       0     5.8    .035       0
#XS Ineff= 2 , 0
               0     110     5.8             110
Permanent Ineff=
       F       F
#Block Obstruct= 2 , 0
                             5.8
Bank Sta=0,5.8
XS Rating Curve= 0
Exp/Cntr=.3,.1

Type RM Length L Ch R = 1 ,2050.00 ,50,50,50
BEGIN DESCRIPTION:
41
END DESCRIPTION:
#Sta/Elev= 10
   -14.5  102.91    -4.5  102.91      -3  104.31       0  104.31     1.6  102.41
     3.2  102.41     5.8  104.91     6.2  104.91     6.4  104.71    16.4  104.71
#Mann= 3 , 0 , 0
   -14.5    .035       0       0    .035       0     5.8    .035       0
#XS Ineff= 2 , 0
               0     110     5.8             110
Permanent Ineff=
       F       F
#Block Obstruct= 2 , 0
                             5.8
Bank Sta=0,5.8
XS Rating Curve= 0
Exp/Cntr=.3,.1

Type RM Length L Ch R = 1 ,2000.00 ,19,19,19
BEGIN DESCRIPTION:
40
END DESCRIPTION:
#Sta/Elev= 11
     -16   102.7      -6   102.7      -3   103.4       0   103.4     1.8   101.6
     3.3   101.6     3.9   102.8     4.9   103.7     5.3   103.7     5.9   103.1
    15.9   103.1
#Mann= 3 , 0 , 0
     -16    .035       0       0    .035       0     4.9    .035       0
#XS Ineff= 2 , 0
               0     110     4.9             110
Permanent Ineff=
       F       F
#Block Obstruct= 2 , 0
                             4.9
Bank Sta=0,4.9
XS Rating Curve= 0
Exp/Cntr=.3,.1

Type RM Length L Ch R = 1 ,1981.00 ,31,31,31
BEGIN DESCRIPTION:
39.031
END DESCRIPTION:
#Sta/Elev= 6
     -10  102.69       0  102.69     2.3  100.89       5  100.89     7.3  102.69
    17.3  102.69
#Mann= 3 , 0 , 0
     -10    .035       0       0    .035       0     7.3    .035       0
#XS Ineff= 2 , 0
               0     110     7.3             110
Permanent Ineff=
       F       F
#Block Obstruct= 2 , 0
                             7.3
Bank Sta=0,7.3
XS Rating Curve= 0
Exp/Cntr=.3,.1

Type RM Length L Ch R = 1 ,1950.00 ,7,7,7
BEGIN DESCRIPTION:
39
END DESCRIPTION:
#Sta/Elev= 14
   -12.2  101.32    -2.2  101.32    -1.2  102.22     -.9  102.22     -.4  102.02
       0  102.02      .3  100.42     2.6  100.42       3  102.02     3.4  102.02
     3.8  102.22     4.4  102.22       5  101.82      15  101.82
#Mann= 3 , 0 , 0
   -12.2    .035       0     2.6    .035       0     3.8    .035       0
#XS Ineff= 2 , 0
             2.6     110     3.8             110
Permanent Ineff=
       F       F
#Block Obstruct= 2 , 0
                             3.8
Bank Sta=2.6,3.8
XS Rating Curve= 0
Exp/Cntr=.3,.1

Type RM Length L Ch R = 1 ,1943.00 ,43,43,43
BEGIN DESCRIPTION:
38.043
END DESCRIPTION:
#Sta/Elev= 14
   -12.2  101.03    -2.2  101.03    -1.2  101.93     -.9  101.93     -.4  101.73
       0  101.73      .3  100.23     2.6  100.23       3  101.73     3.4  101.73
     3.8  101.93     4.4  101.93       5  101.53      15  101.53
#Mann= 3 , 0 , 0
   -12.2    .035       0     2.6    .035       0     3.8    .035       0
#XS Ineff= 2 , 0
             2.6     110     3.8             110
Permanent Ineff=
       F       F
#Block Obstruct= 2 , 0
                             3.8
Bank Sta=2.6,3.8
XS Rating Curve= 0
Exp/Cntr=.3,.1

Type RM Length L Ch R = 1 ,1900.00 ,50,50,50
BEGIN DESCRIPTION:
38
END DESCRIPTION:
#Sta/Elev= 12
   -11.1  101.37    -1.1  101.37     -.7  101.67       0  101.67     1.8  100.07
     2.8  100.07     3.5  100.67     4.4  100.67     6.4  101.67     6.7  101.67
     6.9  101.47    16.9  101.47
#Mann= 3 , 0 , 0
   -11.1    .035       0       0    .035       0     6.4    .035       0
#XS Ineff= 2 , 0
               0     110     6.4             110
Permanent Ineff=
       F       F
#Block Obstruct= 2 , 0
                             6.4
Bank Sta=0,6.4
XS Rating Curve= 0
Exp/Cntr=.3,.1

Type RM Length L Ch R = 1 ,1850.00 ,13,13,13
BEGIN DESCRIPTION:
37
END DESCRIPTION:
#Sta/Elev= 7
     -10   101.7       0   101.7      .2   101.2     2.2    99.8     4.5    99.8
     6.6   101.7    16.6   101.7
#Mann= 3 , 0 , 0
     -10    .035       0       0    .035       0     6.6    .035       0
#XS Ineff= 2 , 0
               0     110     6.6             110
Permanent Ineff=
       F       F
#Block Obstruct= 2 , 0
                             6.6
Bank Sta=0,6.6
XS Rating Curve= 0
Exp/Cntr=.3,.1

Type RM Length L Ch R = 1 ,1837.00 ,37,37,37
BEGIN DESCRIPTION:
36.037
END DESCRIPTION:
#Sta/Elev= 7
     -10  101.82       0  101.82      .2  100.52     2.2   99.12     4.5   99.12
     6.6  101.82    16.6  101.82
#Mann= 3 , 0 , 0
     -10    .035       0       0    .035       0     6.6    .035       0
#XS Ineff= 2 , 0
               0     110     6.6             110
Permanent Ineff=
       F       F
#Block Obstruct= 2 , 0
                             6.6
Bank Sta=0,6.6
XS Rating Curve= 0
Exp/Cntr=.3,.1

Type RM Length L Ch R = 1 ,1800.00 ,50,50,50
BEGIN DESCRIPTION:
36
END DESCRIPTION:
#Sta/Elev= 11
   -10.6   99.84     -.6   99.84     -.4  100.04       0  100.04     2.3   98.54
       4   98.54     4.6   99.34     6.1  100.34     6.3  100.34     6.5  100.14
    16.5  100.14
#Mann= 3 , 0 , 0
   -10.6    .035       0       0    .035       0     6.1    .035       0
#XS Ineff= 2 , 0
               0     105     6.1             105
Permanent Ineff=
       F       F
#Block Obstruct= 2 , 0
                             6.1
Bank Sta=0,6.1
XS Rating Curve= 0
Exp/Cntr=.3,.1

Type RM Length L Ch R = 1 ,1750.00 ,50,50,50
BEGIN DESCRIPTION:
35
END DESCRIPTION:
#Sta/Elev= 11
   -10.6   98.93     -.6   98.93     -.4   99.13       0   99.13     2.3   97.73
       4   97.73     4.6   98.43     6.1   99.43     6.3   99.43     6.5   99.23
    16.5   99.23
#Mann= 3 , 0 , 0
   -10.6    .035       0       0    .035       0     6.1    .035       0
#XS Ineff= 2 , 0
               0     105     6.1             105
Permanent Ineff=
       F       F
#Block Obstruct= 2 , 0
                             6.1
Bank Sta=0,6.1
XS Rating Curve= 0
Exp/Cntr=.3,.1

Type RM Length L Ch R = 1 ,1700.00 ,50,50,50
BEGIN DESCRIPTION:
34
END DESCRIPTION:
#Sta/Elev= 13
   -10.9   98.71     -.9   98.71     -.6   99.01       0   99.01     1.6   97.71
     1.9   97.21     2.7   97.21     2.9   97.81     4.1   97.81     5.9   99.11
     6.5   99.11     6.8   98.81    16.8   98.81
#Mann= 3 , 0 , 0
   -10.9    .035       0       0    .035       0     5.9    .035       0
#XS Ineff= 2 , 0
               0     105     5.9             105
Permanent Ineff=
       F       F
#Block Obstruct= 2 , 0
                             5.9
Bank Sta=0,5.9
XS Rating Curve= 0
Exp/Cntr=.3,.1

Type RM Length L Ch R = 1 ,1650.00 ,7,7,7
BEGIN DESCRIPTION:
33
END DESCRIPTION:
#Sta/Elev= 7
     -10   98.97       0   98.97     2.1   96.57     3.9   96.27     5.6   96.27
     7.8   98.97    17.8   98.97
#Mann= 3 , 0 , 0
     -10    .035       0       0    .035       0     7.8    .035       0
#XS Ineff= 2 , 0
               0     105     7.8             105
Permanent Ineff=
       F       F
#Block Obstruct= 2 , 0
                             7.8
Bank Sta=0,7.8
XS Rating Curve= 0
Exp/Cntr=.3,.1

Type RM Length L Ch R = 1 ,1643.00 ,43,43,43
BEGIN DESCRIPTION:
32.043
END DESCRIPTION:
#Sta/Elev= 7
     -10   99.21       0   99.21     2.1   96.81     3.9   96.51     5.6   96.51
     7.8   99.21    17.8   99.21
#Mann= 3 , 0 , 0
     -10    .035       0       0    .035       0     7.8    .035       0
#XS Ineff= 2 , 0
               0     105     7.8             105
Permanent Ineff=
       F       F
#Block Obstruct= 2 , 0
                             7.8
Bank Sta=0,7.8
XS Rating Curve= 0
Exp/Cntr=.3,.1

Type RM Length L Ch R = 1 ,1600.00 ,8,8,8
BEGIN DESCRIPTION:
32
END DESCRIPTION:
#Sta/Elev= 11
   -11.6    97.4    -1.6    97.4     -.3    98.4       0    98.4     2.7    96.7
     3.3      96     5.1      96     8.4    98.4     9.1    98.4     9.3    98.2
    19.3    98.2
#Mann= 3 , 0 , 0
   -11.6    .035       0       0    .035       0     8.4    .035       0
#XS Ineff= 2 , 0
               0     105     8.4             105
Permanent Ineff=
       F       F
#Block Obstruct= 2 , 0
                             8.4
Bank Sta=0,8.4
XS Rating Curve= 0
Exp/Cntr=.3,.1

Type RM Length L Ch R = 1 ,1592.00 ,42,42,42
BEGIN DESCRIPTION:
31.042
END DESCRIPTION:
#Sta/Elev= 16
   -11.5   97.12    -1.5   97.12    -1.1   97.52     -.8   97.52     -.8   97.72
       0   97.72     1.2   97.22     1.2   96.22       3   96.22       3   97.22
     4.2   97.72       5   97.72     6.3   98.32     7.5   98.32     7.7   98.12
    17.7   98.12
#Mann= 3 , 0 , 0
   -11.5    .035       0       0    .035       0     6.3    .035       0
#XS Ineff= 2 , 0
               0     105     6.3             105
Permanent Ineff=
       F       F
#Block Obstruct= 2 , 0
                             6.3
Bank Sta=0,6.3
XS Rating Curve= 0
Exp/Cntr=.3,.1

Type RM Length L Ch R = 1 ,1550.00 ,50,50,50
BEGIN DESCRIPTION:
31
END DESCRIPTION:
#Sta/Elev= 10
   -10.7   96.63     -.7   96.63     -.5   96.83       0   96.83     2.7   94.83
     5.3   94.83     6.2   97.13     6.8   97.13       7   96.93      17   96.93
#Mann= 3 , 0 , 0
   -10.7    .035       0       0    .035       0       7    .035       0
#XS Ineff= 2 , 0
               0     105       7             105
Permanent Ineff=
       F       F
#Block Obstruct= 2 , 0
                               7
Bank Sta=0,7
XS Rating Curve= 0
Exp/Cntr=.3,.1

Type RM Length L Ch R = 1 ,1500.00 ,50,50,50
BEGIN DESCRIPTION:
30
END DESCRIPTION:
#Sta/Elev= 10
   -10.7    95.7     -.7    95.7     -.5    95.9       0    95.9     2.7    94.4
     5.3    94.4     6.2    96.2     6.8    96.2       7      96      17      96
#Mann= 3 , 0 , 0
   -10.7    .035       0       0    .035       0     6.2    .035       0
#XS Ineff= 2 , 0
               0     100     6.2             100
Permanent Ineff=
       F       F
#Block Obstruct= 2 , 0
                             6.2
Bank Sta=0,6.2
XS Rating Curve= 0
Exp/Cntr=.3,.1

Type RM Length L Ch R = 1 ,1450.00 ,50,50,50
BEGIN DESCRIPTION:
29
END DESCRIPTION:
#Sta/Elev= 7
     -10   96.58       0   96.58     1.2   94.18     2.9   93.78     7.1   93.78
     9.1   96.58    19.1   96.58
#Mann= 3 , 0 , 0
     -10    .035       0       0    .035       0     9.1    .035       0
#XS Ineff= 2 , 0
               0     100     9.1             100
Permanent Ineff=
       F       F
#Block Obstruct= 2 , 0
                             9.1
Bank Sta=0,9.1
XS Rating Curve= 0
Exp/Cntr=.3,.1

Type RM Length L Ch R = 1 ,1400.00 ,50,50,50
BEGIN DESCRIPTION:
28
END DESCRIPTION:
#Sta/Elev= 14
   -10.6    95.2     -.6    95.2     -.3    95.5       0    95.5     2.5    93.7
       3    93.7     3.2    93.2     4.1    93.2     4.3    93.6     5.6    93.6
     8.4    95.4     9.4    95.4      10    94.8      20    94.8
#Mann= 3 , 0 , 0
   -10.6    .035       0       0    .035       0     8.4    .035       0
#XS Ineff= 2 , 0
               0     100     8.4             100
Permanent Ineff=
       F       F
#Block Obstruct= 2 , 0
                             8.4
Bank Sta=0,8.4
XS Rating Curve= 0
Exp/Cntr=.3,.1

Type RM Length L Ch R = 1 ,1350.00 ,50,50,50
BEGIN DESCRIPTION:
27
END DESCRIPTION:
#Sta/Elev= 14
   -10.6   94.74     -.6   94.74     -.3   95.04       0   95.04     2.5   93.34
       3   93.34     3.2   92.84     4.1   92.84     4.3   93.24     5.6   93.24
     8.4   94.94     9.4   94.94      10   94.34      20   94.34
#Mann= 3 , 0 , 0
   -10.6    .035       0       0    .035       0     8.4    .035       0
#XS Ineff= 2 , 0
               0     100     8.4             100
Permanent Ineff=
       F       F
#Block Obstruct= 2 , 0
                             8.4
Bank Sta=0,8.4
XS Rating Curve= 0
Exp/Cntr=.3,.1

Type RM Length L Ch R = 1 ,1300.00 ,50,50,50
BEGIN DESCRIPTION:
26
END DESCRIPTION:
#Sta/Elev= 11
     -16   99.25     -13   97.85     -10   96.45      -7   95.05       0   95.05
       3   92.65       5   92.65     8.6   94.55     9.2   94.55     9.9   94.05
    19.9   94.05
#Mann= 3 , 0 , 0
     -16    .035       0       0    .035       0     8.6    .035       0
#XS Ineff= 2 , 0
               0     100     8.6             100
Permanent Ineff=
       F       F
#Block Obstruct= 2 , 0
                             8.6
Bank Sta=0,8.6
XS Rating Curve= 0
Exp/Cntr=.3,.1

Type RM Length L Ch R = 1 ,1250.00 ,50,50,50
BEGIN DESCRIPTION:
25
END DESCRIPTION:
#Sta/Elev= 12
    -7.5   98.97    -4.5   96.97    -1.5   94.97       0   94.27     1.5   93.37
     2.8   92.07     5.8   92.07       7   93.77     7.3   94.27     8.3   94.27
     9.3   93.47    19.3   93.47
#Mann= 3 , 0 , 0
    -7.5    .035       0       0    .035       0     7.3    .035       0
#XS Ineff= 2 , 0
               0     100     7.3             100
Permanent Ineff=
       F       F
#Block Obstruct= 2 , 0
                             7.3
Bank Sta=0,7.3
XS Rating Curve= 0
Exp/Cntr=.3,.1

Type RM Length L Ch R = 1 ,1200.00 ,50,50,50
BEGIN DESCRIPTION:
24
END DESCRIPTION:
#Sta/Elev= 12
    -7.5   98.34    -4.5   96.34    -1.5   94.34       0   93.94     1.5   92.94
     2.8   91.64     5.8   91.64       7   93.34     7.3   93.64     8.3   93.64
     9.3   92.84    19.3   92.84
#Mann= 3 , 0 , 0
    -7.5    .035       0       0    .035       0     7.3    .035       0
#XS Ineff= 2 , 0
               0     100     7.3             100
Permanent Ineff=
       F       F
#Block Obstruct= 2 , 0
                             7.3
Bank Sta=0,7.3
XS Rating Curve= 0
Exp/Cntr=.3,.1

Type RM Length L Ch R = 1 ,1150.00 ,3,3,3
BEGIN DESCRIPTION:
23
END DESCRIPTION:
#Sta/Elev= 12
    -7.5   98.12    -4.5   96.12    -1.5   94.12       0   93.42     1.5   92.72
     2.8   91.22     5.8   91.22       7   93.12     7.3   93.42     8.3   93.42
     9.3   92.62    19.3   92.62
#Mann= 3 , 0 , 0
    -7.5    .035       0       0    .035       0     7.3    .035       0
#XS Ineff= 2 , 0
               0     100     7.3             100
Permanent Ineff=
       F       F
#Block Obstruct= 2 , 0
                             7.3
Bank Sta=0,7.3
XS Rating Curve= 0
Exp/Cntr=.3,.1

Type RM Length L Ch R = 1 ,1147.00 ,47,47,47
BEGIN DESCRIPTION:
22.047
END DESCRIPTION:
#Sta/Elev= 16
   -12.8   92.52    -2.8   92.52      -2   93.22       0   93.22      .5   91.72
     1.1   91.12     1.6   91.12     2.7   91.12     4.3   91.62     5.8   91.62
     6.3   93.02     6.8   93.02     7.7   93.42     8.6   93.42       9   93.12
      19   93.12
#Mann= 3 , 0 , 0
   -12.8    .035       0       0    .035       0     7.7    .035       0
#XS Ineff= 2 , 0
               0     100     7.7             100
Permanent Ineff=
       F       F
#Block Obstruct= 2 , 0
                             7.7
Bank Sta=0,7.7
XS Rating Curve= 0
Exp/Cntr=.3,.1

Type RM Length L Ch R = 1 ,1100.00 ,50,50,50
BEGIN DESCRIPTION:
22
END DESCRIPTION:
#Sta/Elev= 16
   -11.9   91.78    -1.9   91.78     -.6   92.88       0   92.88      .4   92.48
      .9   92.48     1.3   91.18     2.3   91.18     2.7   90.88     5.1   90.88
     6.3   91.18     6.7   92.48     7.3   92.88     7.9   92.88     8.5   92.28
    18.5   92.28
#Mann= 3 , 0 , 0
   -11.9    .035       0       0    .035       0     7.3    .035       0
#XS Ineff= 2 , 0
               0     100     7.3             100
Permanent Ineff=
       F       F
#Block Obstruct= 2 , 0
                             7.3
Bank Sta=0,7.3
XS Rating Curve= 0
Exp/Cntr=.3,.1

Type RM Length L Ch R = 1 ,1050.00 ,28,28,28
BEGIN DESCRIPTION:
21
END DESCRIPTION:
#Sta/Elev= 7
     -10   92.42       0   92.42     1.2   90.72     2.9   90.32     5.8   90.32
     7.4   92.32    17.4   92.32
#Mann= 3 , 0 , 0
     -10    .035       0       0    .035       0     7.4    .035       0
#XS Ineff= 2 , 0
               0     100     7.4             100
Permanent Ineff=
       F       F
#Block Obstruct= 2 , 0
                             7.4
Bank Sta=0,7.4
XS Rating Curve= 0
Exp/Cntr=.3,.1

Type RM Length L Ch R = 1 ,1022.00 ,22,22,22
BEGIN DESCRIPTION:
20.022
END DESCRIPTION:
#Sta/Elev= 7
     -10   92.26       0   92.26     1.2   90.56     2.9   90.16     5.8   90.16
     7.4   92.16    17.4   92.16
#Mann= 3 , 0 , 0
     -10    .035       0       0    .035       0     7.4    .035       0
#XS Ineff= 2 , 0
               0     100     7.4             100
Permanent Ineff=
       F       F
#Block Obstruct= 2 , 0
                             7.4
Bank Sta=0,7.4
XS Rating Curve= 0
Exp/Cntr=.3,.1

Type RM Length L Ch R = 1 ,1000.00 ,50,50,50
BEGIN DESCRIPTION:
20
END DESCRIPTION:
#Sta/Elev= 12
   -12.5      90    -2.5      90     -.8    91.4       0    91.4     2.1    90.1
     3.4    90.1     3.8    89.8       5    89.8     7.5    91.2       8    91.2
     8.3      91    18.3      91
#Mann= 3 , 0 , 0
   -12.5    .035       0       0    .035       0     7.5    .035       0
#XS Ineff= 2 , 0
               0     100     7.5             100
Permanent Ineff=
       F       F
#Block Obstruct= 2 , 0
                             7.5
Bank Sta=0,7.5
XS Rating Curve= 0
Exp/Cntr=.3,.1

Type RM Length L Ch R = 1 ,950.00  ,25,25,25
BEGIN DESCRIPTION:
19
END DESCRIPTION:
#Sta/Elev= 12
   -12.5      90    -2.5      90     -.8    91.4       0    91.4     2.1    89.9
     3.4    89.9     3.8    89.6       5    89.6     7.5    91.2       8    91.2
     8.3      91    18.3      91
#Mann= 3 , 0 , 0
   -12.5    .035       0       0    .035       0     7.5    .035       0
#XS Ineff= 2 , 0
               0     100     7.5             100
Permanent Ineff=
       F       F
#Block Obstruct= 2 , 0
                             7.5
Bank Sta=0,7.5
XS Rating Curve= 0
Exp/Cntr=.3,.1

Type RM Length L Ch R = 1 ,925.00  ,14,14,14
BEGIN DESCRIPTION:
18.025
END DESCRIPTION:
#Sta/Elev= 9
     -10   90.68       0   90.68      .5   89.38     3.1   89.38     3.6   90.78
       4   91.18     4.6   91.18     5.1   90.68    15.1   90.68
#Mann= 3 , 0 , 0
     -10    .035       0       0    .035       0       4    .035       0
#XS Ineff= 2 , 0
               0     100       4             100
Permanent Ineff=
       F       F
#Block Obstruct= 2 , 0
                               4
Bank Sta=0,4
XS Rating Curve= 0
Exp/Cntr=.3,.1

Type RM Length L Ch R = 1 ,911.00  ,1,1,1
BEGIN DESCRIPTION:
18.011
END DESCRIPTION:
#Sta/Elev= 15
   -18.9   89.45    -8.9   89.45    -7.7   90.15      -2   90.15    -1.1   90.85
       0   90.85      .2   90.15      .2   89.55     4.2   89.55     4.2   90.15
     7.2   90.45     8.1   90.85     8.7   90.85       9   90.55      19   90.55
#Mann= 3 , 0 , 0
   -18.9    .035       0       0    .035       0     8.1    .035       0
#XS Ineff= 2 , 0
               0     100     8.1             100
Permanent Ineff=
       F       F
#Block Obstruct= 2 , 0
                             8.1
Bank Sta=0,8.1
XS Rating Curve= 0
Exp/Cntr=.3,.1

Type RM Length L Ch R = 1 ,910.00  ,10,10,10
BEGIN DESCRIPTION:
18.01
END DESCRIPTION:
#Sta/Elev= 16
   -18.9   89.45    -8.9   89.45    -7.7   90.15      -2   90.15    -1.1   90.85
       0   90.85      .2   90.15      .2   89.55     4.2   88.05     4.2   89.55
     4.2   90.15     7.2   90.45     8.1   90.85     8.7   90.85       9   90.55
      19   90.55
#Mann= 3 , 0 , 0
   -18.9    .035       0       0    .035       0     8.1    .035       0
#XS Ineff= 2 , 0
               0     100     8.1             100
Permanent Ineff=
       F       F
#Block Obstruct= 2 , 0
                             8.1
Bank Sta=0,8.1
XS Rating Curve= 0
Exp/Cntr=.3,.1

Type RM Length L Ch R = 1 ,900.00  ,50,50,50
BEGIN DESCRIPTION:
18
END DESCRIPTION:
#Sta/Elev= 12
   -16.2    89.2    -6.2    89.2    -5.2      90    -1.7      90    -1.2    90.3
       0    90.3      .2    88.2     4.9    88.2     8.1    90.3     8.4    90.3
     8.6    90.1    18.6    90.1
#Mann= 3 , 0 , 0
   -16.2    .035       0       0    .035       0     8.1    .035       0
#XS Ineff= 2 , 0
               0     100     8.1             100
Permanent Ineff=
       F       F
#Block Obstruct= 2 , 0
                             8.1
Bank Sta=0,8.1
XS Rating Curve= 0
Exp/Cntr=.3,.1

Type RM Length L Ch R = 1 ,850.00  ,50,50,50
BEGIN DESCRIPTION:
17
END DESCRIPTION:
#Sta/Elev= 12
   -16.2   88.82    -6.2   88.82    -5.2   89.62    -1.7   89.62    -1.2   89.92
       0   89.92      .2   87.42     4.9   87.42     8.1   89.92     8.4   89.92
     8.6   89.72    18.6   89.72
#Mann= 3 , 0 , 0
   -16.2    .035       0       0    .035       0     8.1    .035       0
#XS Ineff= 2 , 0
               0     100     8.1             100
Permanent Ineff=
       F       F
#Block Obstruct= 2 , 0
                             8.1
Bank Sta=0,8.1
XS Rating Curve= 0
Exp/Cntr=.3,.1

Type RM Length L Ch R = 1 ,800.00  ,50,50,50
BEGIN DESCRIPTION:
16
END DESCRIPTION:
#Sta/Elev= 13
   -15.2   89.53    -5.2   89.53    -4.6   89.83    -4.3   89.83    -3.5   89.43
       0   89.43     3.8   86.83     6.8   86.83     9.2   87.83      12   89.53
    12.7   89.53    13.7   88.53    23.7   88.53
#Mann= 3 , 0 , 0
   -15.2    .035       0       0    .035       0      12    .035       0
#XS Ineff= 2 , 0
               0     100      12             100
Permanent Ineff=
       F       F
#Block Obstruct= 2 , 0
                              12
Bank Sta=0,12
XS Rating Curve= 0
Exp/Cntr=.3,.1

Type RM Length L Ch R = 1 ,750.00  ,50,50,50
BEGIN DESCRIPTION:
15
END DESCRIPTION:
#Sta/Elev= 13
   -15.2   89.34    -5.2   89.34    -4.6   89.64    -4.3   89.64    -3.5   89.24
       0   89.24     3.8   86.44     6.8   86.44     9.2   87.84      12   89.54
    12.7   89.54    13.7   88.54    23.7   88.54
#Mann= 3 , 0 , 0
   -15.2    .035       0       0    .035       0      12    .035       0
#XS Ineff= 2 , 0
               0     100      12             100
Permanent Ineff=
       F       F
#Block Obstruct= 2 , 0
                              12
Bank Sta=0,12
XS Rating Curve= 0
Exp/Cntr=.3,.1

Type RM Length L Ch R = 1 ,700.00  ,13,13,13
BEGIN DESCRIPTION:
14
END DESCRIPTION:
#Sta/Elev= 14
   -14.7   88.69    -4.7   88.69    -4.3   89.09    -3.9   89.09      -3   88.59
       0   88.59     4.5   86.49     7.3   86.49     7.9   86.09    10.4   86.09
    13.2   87.79    13.8   87.79    14.3   87.29    24.3   87.29
#Mann= 3 , 0 , 0
   -14.7    .035       0       0    .035       0    13.2    .035       0
#XS Ineff= 2 , 0
               0     100    13.2             100
Permanent Ineff=
       F       F
#Block Obstruct= 2 , 0
                            13.2
Bank Sta=0,13.2
XS Rating Curve= 0
Exp/Cntr=.3,.1

Type RM Length L Ch R = 1 ,687.00  ,1,1,1
BEGIN DESCRIPTION:
13.037
END DESCRIPTION:
#Sta/Elev= 14
   -14.8   88.71    -4.8   88.71    -4.5   89.11    -4.2   89.11    -3.5   88.61
       0   88.61     2.3   87.31     5.1   86.31     9.1   86.31    11.1   87.31
    12.3   87.91    12.9   87.91    13.4   87.41    23.4   87.41
#Mann= 3 , 0 , 0
   -14.8    .035       0       0    .035       0    12.3    .035       0
#XS Ineff= 2 , 0
               0     100    12.3             100
Permanent Ineff=
       F       F
#Block Obstruct= 2 , 0
                            12.3
Bank Sta=0,12.3
XS Rating Curve= 0
Exp/Cntr=.3,.1

Type RM Length L Ch R = 1 ,686.00  ,36,36,36
BEGIN DESCRIPTION:
13.036
END DESCRIPTION:
#Sta/Elev= 16
   -14.8   88.71    -4.8   88.71    -4.5   89.11    -4.2   89.11    -3.5   88.61
       0   88.61     2.3   87.31     5.1   86.31     5.1   84.81     9.1   84.81
     9.1   86.31    11.9   87.31    13.1   87.91    13.7   87.91    14.2   87.41
    24.2   87.41
#Mann= 3 , 0 , 0
   -14.8    .035       0       0    .035       0    13.1    .035       0
#XS Ineff= 2 , 0
               0     100    13.1             100
Permanent Ineff=
       F       F
#Block Obstruct= 2 , 0
                            13.1
Bank Sta=0,13.1
XS Rating Curve= 0
Exp/Cntr=.3,.1

Type RM Length L Ch R = 1 ,650.00  ,11,11,11
BEGIN DESCRIPTION:
13
END DESCRIPTION:
#Sta/Elev= 14
   -14.8   87.79    -4.8   87.79    -4.5   88.19    -4.2   88.19    -3.5   87.69
       0   87.69     2.3   86.39     5.1   84.89     9.1   84.89    11.9   86.39
    13.1   86.99    13.7   86.99    14.2   86.49    24.2   86.49
#Mann= 3 , 0 , 0
   -14.8    .035       0       0    .035       0    13.1    .035       0
#XS Ineff= 2 , 0
               0     100    13.1             100
Permanent Ineff=
       F       F
#Block Obstruct= 2 , 0
                            13.1
Bank Sta=0,13.1
XS Rating Curve= 0
Exp/Cntr=.3,.1

Type RM Length L Ch R = 1 ,639.00  ,39,39,39
BEGIN DESCRIPTION:
12.039
END DESCRIPTION:
#Sta/Elev= 8
      -9    88.4      -6    87.9      -3    87.4       0    87.4       0    85.1
     4.8    85.1     4.8    87.4    14.8    87.4
#Mann= 3 , 0 , 0
      -9    .035       0       0    .035       0     4.8    .035       0
#XS Ineff= 2 , 0
               0     100     4.8             100
Permanent Ineff=
       F       F
#Block Obstruct= 2 , 0
                             4.8
Bank Sta=0,4.8
XS Rating Curve= 0
Exp/Cntr=.3,.1

Type RM Length L Ch R = 1 ,600.00  ,50,50,50
BEGIN DESCRIPTION:
12
END DESCRIPTION:
#Sta/Elev= 12
   -15.8   87.96    -5.8   87.96    -5.5   88.26    -5.2   88.26      -4   87.26
       0   87.26     2.1   86.26     4.2   85.06     5.2   85.06     5.8   84.56
    10.1   84.56    13.7   86.26
#Mann= 3 , 0 , 0
   -15.8    .035       0       0    .035       0    13.7    .035       0
#XS Ineff= 2 , 0
       0       0     100    13.7       0     100
Permanent Ineff=
       F       F
#Block Obstruct= 2 , 0
                            13.7
Bank Sta=0,13.7
XS Rating Curve= 0
Exp/Cntr=.3,.1

Type RM Length L Ch R = 1 ,550.00  ,20,20,20
BEGIN DESCRIPTION:
11
END DESCRIPTION:
#Sta/Elev= 15
   -15.8   87.39    -5.8   87.39    -5.5   87.69    -5.2   87.69      -4   86.69
       0   86.69     2.1   85.69     4.2   84.89     5.2   84.89     5.8   84.39
    10.1   84.39    13.7   85.69    14.7   85.69    15.9   84.69    25.9   84.69
#Mann= 3 , 0 , 0
   -15.8    .035       0       0    .035       0    13.7    .035       0
#XS Ineff= 2 , 0
               0     100    13.7             100
Permanent Ineff=
       F       F
#Block Obstruct= 2 , 0
                            13.7
Bank Sta=0,13.7
XS Rating Curve= 0
Exp/Cntr=.3,.1

Type RM Length L Ch R = 1 ,530.00  ,20,20,20
BEGIN DESCRIPTION:
10.03
END DESCRIPTION:
#Sta/Elev= 6
     -10   86.53       0   86.53       0   84.43     4.8   84.43     4.8   86.53
    14.8   86.53
#Mann= 3 , 0 , 0
     -10    .035       0       0    .035       0     4.8    .035       0
#XS Ineff= 2 , 0
               0     100     4.8             100
Permanent Ineff=
       F       F
#Block Obstruct= 2 , 0
                             4.8
Bank Sta=0,4.8
XS Rating Curve= 0
Exp/Cntr=.3,.1

Type RM Length L Ch R = 1 ,510.00  ,1,1,1
BEGIN DESCRIPTION:
10.01
END DESCRIPTION:
#Sta/Elev= 19
   -17.1   87.71    -7.1   87.71    -6.8   88.01    -6.3   88.01      -5   87.01
    -4.4   87.01    -1.4   87.01       0   87.01     2.3   85.71     4.9   84.71
     6.3   84.71     6.3   84.51     7.3   84.51     7.3   84.71     9.3   84.71
      12   85.71    12.8   85.71    14.7   84.01    24.7   84.01
#Mann= 3 , 0 , 0
   -17.1    .035       0       0    .035       0      12    .035       0
#XS Ineff= 2 , 0
               0     100      12             100
Permanent Ineff=
       F       F
#Block Obstruct= 2 , 0
                              12
Bank Sta=0,12
XS Rating Curve= 0
Exp/Cntr=.3,.1

Type RM Length L Ch R = 1 ,509.00  ,9,9,9
BEGIN DESCRIPTION:
10.009
END DESCRIPTION:
#Sta/Elev= 17
   -17.1   87.71    -7.1   87.71    -6.8   88.01    -6.3   88.01      -5   87.01
    -4.4   87.01    -1.4   87.01       0   87.01     2.3   85.71     4.9   84.51
     4.9   83.01     9.3   83.01     9.3   84.51      12   85.71    12.8   85.71
    14.7   84.01    24.7   84.01
#Mann= 3 , 0 , 0
   -17.1    .035       0       0    .035       0      12    .035       0
#XS Ineff= 2 , 0
               0     100      12             100
Permanent Ineff=
       F       F
#Block Obstruct= 2 , 0
                              12
Bank Sta=0,12
XS Rating Curve= 0
Exp/Cntr=.3,.1

Type RM Length L Ch R = 1 ,500.00  ,50,50,50
BEGIN DESCRIPTION:
10
END DESCRIPTION:
#Sta/Elev= 11
    -6.6   86.86    -1.6   86.86       0   86.86       3   85.06     3.7   84.66
     5.7   83.36     9.7   83.36    13.2   85.36      14   85.36    15.5   84.06
    25.5   84.06
#Mann= 3 , 0 , 0
    -6.6    .035       0       0    .035       0    13.2    .035       0
#XS Ineff= 2 , 0
               0      95    13.2              95
Permanent Ineff=
       F       F
#Block Obstruct= 2 , 0
                            13.2
Bank Sta=0,13.2
XS Rating Curve= 0
Exp/Cntr=.3,.1

Type RM Length L Ch R = 1 ,450.00  ,50,50,50
BEGIN DESCRIPTION:
9
END DESCRIPTION:
#Sta/Elev= 11
    -6.6   85.52    -1.6   85.52       0   85.52       3   83.72     3.7   83.32
     5.7   82.92     9.7   82.92    13.2   84.92      14   84.92    15.5   83.62
    25.5   83.62
#Mann= 3 , 0 , 0
    -6.6    .035       0       0    .035       0    13.2    .035       0
#XS Ineff= 2 , 0
               0      95    13.2              95
Permanent Ineff=
       F       F
#Block Obstruct= 2 , 0
                            13.2
Bank Sta=0,13.2
XS Rating Curve= 0
Exp/Cntr=.3,.1

Type RM Length L Ch R = 1 ,400.00  ,18,18,18
BEGIN DESCRIPTION:
8
END DESCRIPTION:
#Sta/Elev= 13
   -14.3   83.86    -4.3   83.86    -3.5   84.56       0   84.56       3   82.96
       4   82.96     4.4   82.56     7.7   82.56     8.2   83.26      11   84.86
    11.4   84.86    11.6   84.66    21.6   84.66
#Mann= 3 , 0 , 0
   -14.3    .035       0       0    .035       0      11    .035       0
#XS Ineff= 2 , 0
               0      90      11              90
Permanent Ineff=
       F       F
#Block Obstruct= 2 , 0
                              11
Bank Sta=0,11
XS Rating Curve= 0
Exp/Cntr=.3,.1

Type RM Length L Ch R = 1 ,382.00  ,1,1,1
BEGIN DESCRIPTION:
7.032
END DESCRIPTION:
#Sta/Elev= 12
     -15   83.38      -5   83.38    -3.5   84.38       0   84.38     2.7   82.88
     4.7   82.88     4.7   82.68     5.6   82.68     5.6   82.88     7.2   82.88
    10.1   84.18    20.1   84.18
#Mann= 3 , 0 , 0
     -15    .035       0       0    .035       0    10.1    .035       0
#XS Ineff= 2 , 0
               0      90    10.1              90
Permanent Ineff=
       F       F
#Block Obstruct= 2 , 0
                            10.1
Bank Sta=0,10.1
XS Rating Curve= 0
Exp/Cntr=.3,.1

Type RM Length L Ch R = 1 ,381.00  ,7,7,7
BEGIN DESCRIPTION:
7.031
END DESCRIPTION:
#Sta/Elev= 10
     -15   83.38      -5   83.38    -3.5   84.38       0   84.38     2.7   82.88
     2.7   81.18     8.2   81.18     8.2   82.88    11.1   84.08    21.1   84.08
#Mann= 3 , 0 , 0
     -15    .035       0       0    .035       0    11.1    .035       0
#XS Ineff= 2 , 0
               0      90    11.1              90
Permanent Ineff=
       F       F
#Block Obstruct= 2 , 0
                            11.1
Bank Sta=0,11.1
XS Rating Curve= 0
Exp/Cntr=.3,.1

Type RM Length L Ch R = 1 ,374.00  ,24,24,24
BEGIN DESCRIPTION:
7.024
END DESCRIPTION:
#Sta/Elev= 10
   -17.8   83.17    -7.8   83.17    -6.5   84.27    -3.5   84.27      -2   83.57
       0   83.57       0   81.37     4.7   81.37     4.7   83.57    14.7   83.57
#Mann= 3 , 0 , 0
   -17.8    .035       0       0    .035       0     4.7    .035       0
#XS Ineff= 2 , 0
               0      90     4.7              90
Permanent Ineff=
       F       F
#Block Obstruct= 2 , 0
                             4.7
Bank Sta=0,4.7
XS Rating Curve= 0
Exp/Cntr=.3,.1

Type RM Length L Ch R = 1 ,350.00  ,50,50,50
BEGIN DESCRIPTION:
7
END DESCRIPTION:
#Sta/Elev= 12
   -13.5   82.95    -3.5   82.95      -3   93.45       0   83.45       0   83.35
     2.1   82.05     4.2   81.15     8.7   81.15    11.9   82.65    12.6   82.65
    13.9   81.55    23.9   81.55
#Mann= 3 , 0 , 0
   -13.5    .035       0       0    .035       0    11.9    .035       0
#XS Ineff= 2 , 0
               0      90    11.9              90
Permanent Ineff=
       F       F
#Block Obstruct= 2 , 0
                            11.9
Bank Sta=0,11.9
XS Rating Curve= 0
Exp/Cntr=.3,.1

Type RM Length L Ch R = 1 ,300.00  ,25,25,25
BEGIN DESCRIPTION:
6
END DESCRIPTION:
#Sta/Elev= 11
   -13.5   82.73    -3.5   82.73       0   83.23       0   83.13     2.1   81.83
     4.2   80.53     8.7   80.53    11.9   82.43    12.6   82.43    13.9   81.33
    23.9   81.33
#Mann= 3 , 0 , 0
   -13.5    .035       0       0    .035       0    11.9    .035       0
#XS Ineff= 2 , 0
               0      90    11.9              90
Permanent Ineff=
       F       F
#Block Obstruct= 2 , 0
                            11.9
Bank Sta=0,11.9
XS Rating Curve= 0
Exp/Cntr=.3,.1

Type RM Length L Ch R = 1 ,275.00  ,25,25,25
BEGIN DESCRIPTION:
5.025
END DESCRIPTION:
#Sta/Elev= 19
   -14.2   81.67    -4.2   81.67      -3   82.57       0   82.57     2.3   81.27
     4.3   80.27     6.1   80.27     6.1   79.77     6.7   79.77     6.7   80.27
     7.6   80.27     7.6   79.77     8.2   79.77     8.2   80.27    10.4   80.27
    13.6   81.97    14.4   81.97    15.2   81.17    25.2   81.17
#Mann= 3 , 0 , 0
   -14.2    .035       0       0    .035       0    13.6    .035       0
#XS Ineff= 2 , 0
               0      90    13.6              90
Permanent Ineff=
       F       F
#Block Obstruct= 2 , 0
                            13.6
Bank Sta=0,13.6
XS Rating Curve= 0
Exp/Cntr=.3,.1

Type RM Length L Ch R = 1 ,250.00  ,50,50,50
BEGIN DESCRIPTION:
5
END DESCRIPTION:
#Sta/Elev= 16
   -15.4   82.61    -5.4   82.61      -5   82.91    -4.6   82.91      -4   82.51
      -3   82.51       0   82.51       3   81.01     5.5   79.81     6.5   79.81
       8   80.31     9.2   80.31    12.2   82.01    12.8   82.01    13.4   81.31
    23.4   81.31
#Mann= 3 , 0 , 0
   -15.4    .035       0       0    .035       0    12.2    .035       0
#XS Ineff= 2 , 0
               0      90    12.2              90
Permanent Ineff=
       F       F
#Block Obstruct= 2 , 0
                            12.2
Bank Sta=0,12.2
XS Rating Curve= 0
Exp/Cntr=.3,.1
