--- MSC.prj (project) ---

Proj Title=MSC
Current Plan=p01
Default Exp/Contr=.3,.1
SI Units
Geom File=g01
Flow File=f01
Plan File=p01
Y Axis Title=Elevation
X Axis Title(PF)=Main Channel Distance
X Axis Title(XS)=Station
BEGIN DESCRIPTION:
           BACK WATER COMPUTATION
      APPLICATION OF HEC-2 BY Samju Construction Engineering
      namshim-cheon: 10,20,30,50,80 yr
END DESCRIPTION:
DSS Export Rating Curves= 0
DSS Export Rating Curve Sorted= 0
DSS Export Volume Flow Curves= 0
DXF OffsetX= 0
DXF OffsetY= 0
DXF ScaleX= 1
DXF ScaleY= 10

--- MSC.p01 (plan) ---

Plan Title=Imported Plan 01
Version=Version 3.0.1  Mar 2001
Short Identifier=Imported Pla
Geom File=g01
Flow File=f01
Subcritical Flow
K Sum by GR= 0
Std Step Tol= 0.003
Critical Tol= 0.003
Num of Std Step Trials= 20
Max Error Tol= 0.1
Flow Tol Ratio= 0.001
Split Flow NTrial= 30
Split Flow Tol= 0.02
Split Flow Ratio= 0.02
Log Output Level= 0
Friction Slope Method= 1
Unsteady Friction Slope Method= 2
Parabolic Critical Depth
Global Vel Dist= 0 , 0 , 0
Global Log Level= 0
CheckData=True
Encroach Param=-1 ,0,0, 0
Computation Interval=1HOUR
Output Interval=1HOUR
Run HTab= 0
Run UNet= 0
Run PostProcess= 0
UNET Theta= 1
UNET ZTol= 0.02
UNET ZSATol= 0.1
UNET MxIter= 20
UNET MaxInSteps= 20
UNET DtIC= 0
UNET DtMin= 0
UNET MaxCRTS= 20
UNET WFStab= 2
UNET SFStab= 1
UNET WFX= 1
UNET SFX= 1
UNET Convert EG Bridges=-1
UNET Use Existing IB Tables=-1
Instantaneous Interval=1HOUR
Write IC File= 0
Write Velocity= 0
Write Detailed= 0

--- MSC.f01 (steady flow) ---

Flow Title=Imported Flow 01
Version=Version 3.0.1  Mar 2001
Number of Profiles= 5
Profile Names=10YR,20YR,30YR,50YR,80YR
River Rch & RM=RIVER-1,Reach-1         ,2099.00
    13.2   14.53    15.3   16.28   17.19
River Rch & RM=RIVER-1,Reach-1         ,1093.00
   27.85   30.68   32.33   34.42   36.34
Boundary for River Rch & Prof#=RIVER-1,Reach-1         , 1
Up Type= 0
Dn Type= 3
Dn Slope=.045
Boundary for River Rch & Prof#=RIVER-1,Reach-1         , 2
Up Type= 0
Dn Type= 3
Dn Slope=.045
Boundary for River Rch & Prof#=RIVER-1,Reach-1         , 3
Up Type= 0
Dn Type= 3
Dn Slope=.045
Boundary for River Rch & Prof#=RIVER-1,Reach-1         , 4
Up Type= 0
Dn Type= 3
Dn Slope=.045
Boundary for River Rch & Prof#=RIVER-1,Reach-1         , 5
Up Type= 0
Dn Type= 3
Dn Slope=.045
DSS Import GetInterval= 0
DSS Import GetPeak= 0
DSS Import FillOption= 0

--- MSC.g01 (geometry) ---

Geom Title=Imported Geom 01
Version=Version 3.0.1  Mar 2001

River Reach=RIVER-1         ,Reach-1
Reach XY= 2
              .5             .95              .5             .05

Type RM Length L Ch R = 1 ,2099.00 ,49,49,49
BEGIN DESCRIPTION:
40.049
END DESCRIPTION:
#Sta/Elev= 10
   -11.8  151.74    -1.8  151.74     -.6  152.94       0  152.94     1.6  151.84
     2.8  151.84     5.8  153.54     8.8  155.04    11.8  156.54    14.3  157.74
#Mann= 3 , 0 , 0
   -11.8    .035       0       0    .035       0     5.8    .035       0
#XS Ineff= 2 , 0
               0  152.94     5.8          153.54
Permanent Ineff=
       F       F
Bank Sta=0,5.8
XS Rating Curve= 0
Exp/Cntr=.3,.1

Type RM Length L Ch R = 1 ,2050.00 ,50,50,50
BEGIN DESCRIPTION:
40
END DESCRIPTION:
#Sta/Elev= 12
   -11.6  147.31    -1.6  147.31     -.8  148.01       0  148.01      .7  147.11
      .8  146.41     2.1  146.41     4.3  148.51     7.3  150.01    10.3  151.51
    12.3  152.71    22.3  152.71
#Mann= 3 , 0 , 0
   -11.6    .035       0       0    .035       0     4.3    .035       0
#XS Ineff= 2 , 0
               0  148.01     4.3          148.51
Permanent Ineff=
       F       F
Bank Sta=0,4.3
XS Rating Curve= 0
Exp/Cntr=.3,.1

Type RM Length L Ch R = 1 ,2000.00 ,50,50,50
BEGIN DESCRIPTION:
39
END DESCRIPTION:
#Sta/Elev= 11
   -14.4  145.05    -4.4  145.05    -3.2  143.85    -1.7  143.85     -.5  144.45
       0  144.45     1.4  142.75     2.4  142.75     4.4  144.25     7.4  146.05
     8.9  147.55
#Mann= 3 , 0 , 0
   -14.4    .035       0       0    .035       0     4.4    .035       0
#XS Ineff= 2 , 0
               0  144.45     4.4          144.25
Permanent Ineff=
       F       F
Bank Sta=0,4.4
XS Rating Curve= 0
Exp/Cntr=.3,.1

Type RM Length L Ch R = 1 ,1950.00 ,28,28,28
BEGIN DESCRIPTION:
38
END DESCRIPTION:
#Sta/Elev= 11
   -14.4  141.49    -4.4  141.49    -3.2  140.29    -1.7  140.29     -.5  140.89
       0  140.89     1.4  139.19     2.4  139.19     4.4  140.69     7.4  142.49
     8.9  143.99
#Mann= 3 , 0 , 0
   -14.4    .035       0       0    .035       0     4.4    .035       0
#XS Ineff= 2 , 0
               0  140.89     4.4          140.69
Permanent Ineff=
       F       F
Bank Sta=0,4.4
XS Rating Curve= 0
Exp/Cntr=.3,.1

Type RM Length L Ch R = 1 ,1922.00 ,6,6,6
BEGIN DESCRIPTION:
37.027
END DESCRIPTION:
#Sta/Elev= 10
     -10  139.75       0  139.75      .3  138.15     1.7  138.15     1.7  138.05
     1.9  138.05     3.5  138.25     3.7  139.65     6.7  139.95     9.7  140.45
#Mann= 3 , 0 , 0
     -10    .035       0       0    .035       0     3.7    .035       0
#XS Ineff= 2 , 0
               0  139.75     3.7          139.65
Permanent Ineff=
       F       F
Bank Sta=0,3.7
XS Rating Curve= 0
Exp/Cntr=.3,.1

Type RM Length L Ch R = 1 ,1916.00 ,1,1,1
BEGIN DESCRIPTION:
37.021
END DESCRIPTION:
#Sta/Elev= 14
     -10  139.23       0  139.23     2.2  138.33     2.9  138.03     3.2  138.03
     3.2  137.73     4.8  137.73     4.8  138.13     5.1  138.13     6.7  138.33
       7  139.43      10  139.73      13  140.23      16  140.73
#Mann= 3 , 0 , 0
     -10    .035       0       0    .035       0       7    .035       0
#XS Ineff= 2 , 0
               0  139.23       7          139.43
Permanent Ineff=
       F       F
Bank Sta=0,7
XS Rating Curve= 0
Exp/Cntr=.3,.1

Type RM Length L Ch R = 1 ,1915.00 ,20,20,20
BEGIN DESCRIPTION:
37.02
END DESCRIPTION:
#Sta/Elev= 14
     -10  139.23       0  139.23     2.2  138.33     2.9  138.03     3.2  138.03
     3.2  137.23     4.8  137.23     4.8  138.03     4.8  138.43     5.1  138.43
     6.7  138.63       7  139.73      10  140.03      13  140.53
#Mann= 3 , 0 , 0
     -10    .035       0       0    .035       0       7    .035       0
#XS Ineff= 2 , 0
               0  139.23       7          139.73
Permanent Ineff=
       F       F
Bank Sta=0,7
XS Rating Curve= 0
Exp/Cntr=.3,.1

Type RM Length L Ch R = 1 ,1895.00 ,50,50,50
BEGIN DESCRIPTION:
37
END DESCRIPTION:
#Sta/Elev= 14
   -12.7  136.41    -2.7  136.41     -.8  138.01       0  138.01     1.4  136.81
     2.4  136.21       4  136.21     4.7  136.31     5.5  136.41     8.5  138.41
    11.5  140.41    11.9  140.41    12.1  140.21    22.1  140.21
#Mann= 3 , 0 , 0
   -12.7    .035       0       0    .035       0     8.5    .035       0
#XS Ineff= 2 , 0
               0  138.01     8.5          138.41
Permanent Ineff=
       F       F
Bank Sta=0,8.5
XS Rating Curve= 0
Exp/Cntr=.3,.1

Type RM Length L Ch R = 1 ,1845.00 ,41,41,41
BEGIN DESCRIPTION:
36
END DESCRIPTION:
#Sta/Elev= 14
   -12.7  134.71    -2.7  134.71     -.8  136.31       0  136.31     1.4  135.01
     2.4   134.3       4  134.31     4.7  134.51     5.5  134.61     8.5  136.61
    11.5  138.61    11.9  138.61    12.1  138.41    22.1  138.41
#Mann= 3 , 0 , 0
   -12.7    .035       0       0    .035       0     8.5    .035       0
#XS Ineff= 2 , 0
               0  136.31     8.5          136.61
Permanent Ineff=
       F       F
Bank Sta=0,8.5
XS Rating Curve= 0
Exp/Cntr=.3,.1

Type RM Length L Ch R = 1 ,1804.00 ,2,2,2
BEGIN DESCRIPTION:
35.01
END DESCRIPTION:
#Sta/Elev= 11
   -11.4  134.65    -1.4  134.65      -1  134.65     -.5  134.65       0  134.35
      .7  133.15     5.6  133.15       6  133.55     7.2  133.75     8.3  134.25
    11.6  134.25
#Mann= 3 , 0 , 0
   -11.4    .035       0      -1    .035       0     8.3    .035       0
#XS Ineff= 2 , 0
              -1  134.65     8.3          134.25
Permanent Ineff=
       F       F
Bank Sta=-1,8.3
XS Rating Curve= 0
Exp/Cntr=.3,.1

Type RM Length L Ch R = 1 ,1802.00 ,1,1,1
BEGIN DESCRIPTION:
35.009
END DESCRIPTION:
#Sta/Elev= 13
   -11.4  134.65    -1.4  134.65      -1  134.65     -.5  134.35       0  134.35
      .7  133.15      .7  132.45     5.6  132.45     5.6  133.15       6  133.55
     7.2  133.75     8.3  134.25    11.6  134.25
#Mann= 3 , 0 , 0
   -11.4    .035       0      -1    .035       0     8.3    .035       0
#XS Ineff= 2 , 0
              -1  134.65     8.3          134.25
Permanent Ineff=
       F       F
Bank Sta=-1,8.3
XS Rating Curve= 0
Exp/Cntr=.3,.1

Type RM Length L Ch R = 1 ,1801.00 ,1,1,1
BEGIN DESCRIPTION:
35.008
END DESCRIPTION:
#Sta/Elev= 11
   -11.4  134.52    -1.4  134.52      -1  134.52     -.5  134.22       0  134.22
      .7  132.42     5.6  132.42       6  133.42     7.2  133.62     8.3  134.12
    11.6  134.12
#Mann= 3 , 0 , 0
   -11.4    .035       0      -1    .035       0     8.3    .035       0
#XS Ineff= 2 , 0
              -1  134.52     8.3          134.12
Permanent Ineff=
       F       F
Bank Sta=-1,8.3
XS Rating Curve= 0
Exp/Cntr=.3,.1

Type RM Length L Ch R = 1 ,1800.00 ,7,7,7
BEGIN DESCRIPTION:
35.007
END DESCRIPTION:
#Sta/Elev= 13
   -11.4  134.52    -1.4  134.52      -1  134.52     -.5  134.22       0  134.22
      .7  132.42      .7  131.72     5.6  131.72     5.6  132.42       6  133.42
     7.2  133.62     8.3  134.12     116  134.12
#Mann= 3 , 0 , 0
   -11.4    .035       0      -1    .035       0     8.3    .035       0
#XS Ineff= 2 , 0
              -1  134.52     8.3          134.12
Permanent Ineff=
       F       F
Bank Sta=-1,8.3
XS Rating Curve= 0
Exp/Cntr=.3,.1

Type RM Length L Ch R = 1 ,1793.00 ,42,42,42
BEGIN DESCRIPTION:
35
END DESCRIPTION:
#Sta/Elev= 9
     -10  134.09       0  134.09      .4  133.59      .5  131.69     3.5  131.69
     3.6  132.79       4  133.09       7  133.39      10  133.79
#Mann= 3 , 0 , 0
     -10    .035       0       0    .035       0       7    .035       0
#XS Ineff= 2 , 0
               0  134.09       7          133.39
Permanent Ineff=
       F       F
Bank Sta=0,7
XS Rating Curve= 0
Exp/Cntr=.3,.1

Type RM Length L Ch R = 1 ,1751.00 ,1,1,1
BEGIN DESCRIPTION:
34.008
END DESCRIPTION:
#Sta/Elev= 10
   -12.9  130.86    -2.9  130.86      -2  131.36       0  131.36       2  130.76
     4.2  130.76     7.2  131.56     7.5  131.56     7.6  131.46    17.6  131.46
#Mann= 3 , 0 , 0
   -12.9    .035       0       0    .035       0     7.2    .035       0
#XS Ineff= 2 , 0
               0  131.36     7.2          131.56
Permanent Ineff=
       F       F
Bank Sta=0,7.2
XS Rating Curve= 0
Exp/Cntr=.3,.1

Type RM Length L Ch R = 1 ,1750.00 ,7,7,7
BEGIN DESCRIPTION:
34.007
END DESCRIPTION:
#Sta/Elev= 12
   -12.9  130.86    -2.9  130.86      -2  131.36       0  131.36       2  130.76
       2  130.06     4.2  130.06     4.2  130.76     7.2  131.56     7.5  131.56
     7.6  131.46    17.6  131.46
#Mann= 3 , 0 , 0
   -12.9    .035       0       0    .035       0     7.2    .035       0
#XS Ineff= 2 , 0
               0  131.36     7.2          131.56
Permanent Ineff=
       F       F
Bank Sta=0,7.2
XS Rating Curve= 0
Exp/Cntr=.3,.1

Type RM Length L Ch R = 1 ,1743.00 ,50,50,50
BEGIN DESCRIPTION:
34
END DESCRIPTION:
#Sta/Elev= 12
   -13.2  130.12    -3.2  130.12    -2.2  131.12       0  131.12      .8  130.62
       2  130.32     2.5  129.92     4.2  129.92     7.2  132.32     7.5  132.32
     7.6  132.22    17.6  132.22
#Mann= 3 , 0 , 0
   -13.2    .035       0       0    .035       0     7.2    .035       0
#XS Ineff= 2 , 0
               0  131.12     7.2          132.32
Permanent Ineff=
       F       F
Bank Sta=0,7.2
XS Rating Curve= 0
Exp/Cntr=.3,.1

Type RM Length L Ch R = 1 ,1693.00 ,5,5,5
BEGIN DESCRIPTION:
33
END DESCRIPTION:
#Sta/Elev= 11
     -10  129.59       0  129.59     1.3  128.49     2.6  128.39     5.6  128.39
       6  128.59     8.2  128.69      10  130.19    12.5  130.19    13.1  129.79
    23.1  129.79
#Mann= 3 , 0 , 0
     -10    .035       0       0    .035       0      10    .035       0
#XS Ineff= 2 , 0
               0  129.59      10          130.19
Permanent Ineff=
       F       F
Bank Sta=0,10
XS Rating Curve= 0
Exp/Cntr=.3,.1

Type RM Length L Ch R = 1 ,1688.00 ,1,1,1
BEGIN DESCRIPTION:
32.045
END DESCRIPTION:
#Sta/Elev= 11
     -10  129.28       0  129.28     1.3  127.58     2.6  127.48     5.6  127.48
       6  127.78     8.2  127.98      10  129.78    12.5  129.78    13.1  129.38
    23.1  129.38
#Mann= 3 , 0 , 0
     -10    .035       0       0    .035       0      10    .035       0
#XS Ineff= 2 , 0
               0  129.28      10          129.78
Permanent Ineff=
       F       F
Bank Sta=0,10
XS Rating Curve= 0
Exp/Cntr=.3,.1

Type RM Length L Ch R = 1 ,1687.00 ,44,44,44
BEGIN DESCRIPTION:
32.044
END DESCRIPTION:
#Sta/Elev= 13
     -10  129.28       0  129.28     1.3  127.58     2.6  127.48     2.6  127.08
     5.6  127.08     5.6  127.48       6  127.78     8.2  127.98      10  129.78
    12.5  129.78    13.1  129.38    23.1  129.38
#Mann= 3 , 0 , 0
     -10    .035       0       0    .035       0      10    .035       0
#XS Ineff= 2 , 0
               0  129.28      10          129.78
Permanent Ineff=
       F       F
Bank Sta=0,10
XS Rating Curve= 0
Exp/Cntr=.3,.1

Type RM Length L Ch R = 1 ,1643.00 ,22,22,22
BEGIN DESCRIPTION:
32
END DESCRIPTION:
#Sta/Elev= 11
   -13.4  127.56    -3.4  127.56    -2.2  128.06       0  128.06     1.5  126.86
     3.8  126.06     5.3  126.06     7.8  128.86    10.3  128.86    10.7  128.56
    20.7  128.56
#Mann= 3 , 0 , 0
   -13.4    .035       0       0    .035       0     7.8    .035       0
#XS Ineff= 2 , 0
               0  128.06     7.8          128.86
Permanent Ineff=
       F       F
Bank Sta=0,7.8
XS Rating Curve= 0
Exp/Cntr=.3,.1

Type RM Length L Ch R = 1 ,1621.00 ,1,1,1
BEGIN DESCRIPTION:
31.028
END DESCRIPTION:
#Sta/Elev= 11
   -13.4  126.11    -3.4  126.11    -2.2  127.31       0  127.31      .4  126.71
     2.7  125.91     4.2  125.91     6.7  128.11     9.2  128.11     9.6  127.81
    19.6  127.81
#Mann= 3 , 0 , 0
   -13.4    .035       0       0    .035       0     6.7    .035       0
#XS Ineff= 2 , 0
               0  127.31     6.7          128.11
Permanent Ineff=
       F       F
Bank Sta=0,6.7
XS Rating Curve= 0
Exp/Cntr=.3,.1

Type RM Length L Ch R = 1 ,1620.00 ,18,18,18
BEGIN DESCRIPTION:
31.027
END DESCRIPTION:
#Sta/Elev= 13
   -13.4  126.11    -3.4  126.11    -2.2  127.31       0  127.31      .4  126.71
     2.7  125.91     2.7  125.31     4.2  125.31     4.2  125.91     6.7  128.11
     9.2  128.11     9.6  127.81    19.6  127.81
#Mann= 3 , 0 , 0
   -13.4    .035       0       0    .035       0     6.7    .035       0
#XS Ineff= 2 , 0
               0  127.31     6.7          128.11
Permanent Ineff=
       F       F
Bank Sta=0,6.7
XS Rating Curve= 0
Exp/Cntr=.3,.1

Type RM Length L Ch R = 1 ,1602.00 ,9,9,9
BEGIN DESCRIPTION:
31.009
END DESCRIPTION:
#Sta/Elev= 11
     -13  126.18      -3  126.18      -2  126.78       0  126.78     1.1  126.38
     2.9  125.38     7.9  125.38     9.9  127.38    12.9  127.38    13.5  126.78
    23.5  126.78
#Mann= 3 , 0 , 0
     -13    .035       0       0    .035       0     9.9    .035       0
#XS Ineff= 2 , 0
               0  126.78     9.9          127.38
Permanent Ineff=
       F       F
Bank Sta=0,9.9
XS Rating Curve= 0
Exp/Cntr=.3,.1

Type RM Length L Ch R = 1 ,1593.00 ,33,33,33
BEGIN DESCRIPTION:
31
END DESCRIPTION:
#Sta/Elev= 11
     -10  126.57       0  126.57       3  125.67     3.8  125.57     5.8  124.27
    10.1  124.27    11.8  124.47    13.8  125.57    15.8  125.57    16.5  125.47
    26.5  125.47
#Mann= 3 , 0 , 0
     -10    .035       0       0    .035       0    13.8    .035       0
#XS Ineff= 2 , 0
               0  126.57    13.8          125.57
Permanent Ineff=
       F       F
Bank Sta=0,13.8
XS Rating Curve= 0
Exp/Cntr=.3,.1

Type RM Length L Ch R = 1 ,1560.00 ,17,17,17
BEGIN DESCRIPTION:
30.017
END DESCRIPTION:
#Sta/Elev= 11
     -10  127.33       0  127.33       3  125.93     3.8  125.83     5.8  123.73
    10.1  123.73    11.8  123.93    13.8  125.03    15.8  125.03    16.5  124.93
    26.5  124.93
#Mann= 3 , 0 , 0
     -10    .035       0       0    .035       0    13.8    .035       0
#XS Ineff= 2 , 0
               0  127.33    13.8          125.03
Permanent Ineff=
       F       F
Bank Sta=0,13.8
XS Rating Curve= 0
Exp/Cntr=.3,.1

Type RM Length L Ch R = 1 ,1543.00 ,35,35,35
BEGIN DESCRIPTION:
30
END DESCRIPTION:
#Sta/Elev= 14
     -12  126.66      -2  126.66    -1.7  126.86       0  126.86       3  124.96
     4.2  124.46     5.9  122.66    10.4  122.66    11.2  123.06    11.6  123.66
    13.7  124.86    15.7  124.86    16.5  124.06    26.5  124.06
#Mann= 3 , 0 , 0
     -12    .035       0       0    .035       0    13.7    .035       0
#XS Ineff= 2 , 0
               0  126.86    13.7          124.86
Permanent Ineff=
       F       F
Bank Sta=0,13.7
XS Rating Curve= 0
Exp/Cntr=.3,.1

Type RM Length L Ch R = 1 ,1508.00 ,15,15,15
BEGIN DESCRIPTION:
29.015
END DESCRIPTION:
#Sta/Elev= 11
   -13.2  124.11    -3.2  124.11    -2.2  125.01       0  125.01     3.2  123.51
     5.2  122.31    10.2  122.31    12.7  123.81    14.9  123.81      17  122.91
      27  122.91
#Mann= 3 , 0 , 0
   -13.2    .035       0       0    .035       0    12.7    .035       0
#XS Ineff= 2 , 0
               0  125.01    12.7          123.81
Permanent Ineff=
       F       F
Bank Sta=0,12.7
XS Rating Curve= 0
Exp/Cntr=.3,.1

Type RM Length L Ch R = 1 ,1493.00 ,34,34,34
BEGIN DESCRIPTION:
29
END DESCRIPTION:
#Sta/Elev= 10
   -13.7     123    -3.7     123    -2.2   124.4       0   124.4     1.8   122.8
       4     121       9     121    11.2   122.9    13.6   122.9    14.8   122.5
#Mann= 3 , 0 , 0
   -13.7    .035       0       0    .035       0    11.2    .035       0
#XS Ineff= 2 , 0
               0   124.4    11.2           122.9
Permanent Ineff=
       F       F
Bank Sta=0,11.2
XS Rating Curve= 0
Exp/Cntr=.3,.1

Type RM Length L Ch R = 1 ,1459.00 ,1,1,1
BEGIN DESCRIPTION:
28.016
END DESCRIPTION:
#Sta/Elev= 11
   -13.7  121.48    -3.7  121.48    -2.2  122.88       0  122.88     1.8  121.68
       4  120.48       9  120.48    11.2  121.48    13.6  121.48    14.8  121.08
    24.8  121.08
#Mann= 3 , 0 , 0
   -13.7    .035       0       0    .035       0    11.2    .035       0
#XS Ineff= 2 , 0
               0  122.88    11.2          121.48
Permanent Ineff=
       F       F
Bank Sta=0,11.2
XS Rating Curve= 0
Exp/Cntr=.3,.1

Type RM Length L Ch R = 1 ,1458.00 ,15,15,15
BEGIN DESCRIPTION:
28.015
END DESCRIPTION:
#Sta/Elev= 13
   -13.7  121.48    -3.7  121.48    -2.2  122.88       0  122.88     1.8  121.68
       4  120.48       4  119.68       9  119.68       9  120.48    11.2  121.48
    13.6  121.48    14.8  121.08    24.8  121.08
#Mann= 3 , 0 , 0
   -13.7    .035       0       0    .035       0    11.2    .035       0
#XS Ineff= 2 , 0
               0  122.88    11.2          121.48
Permanent Ineff=
       F       F
Bank Sta=0,11.2
XS Rating Curve= 0
Exp/Cntr=.3,.1

Type RM Length L Ch R = 1 ,1443.00 ,34,34,34
BEGIN DESCRIPTION:
28
END DESCRIPTION:
#Sta/Elev= 13
   -12.9  121.23    -2.9  121.23    -2.2  121.93       0  121.93       3  120.13
       5  119.83     5.8  119.83     7.8  120.23     8.9  120.53      11  121.83
    13.3  121.83    14.3  121.03    24.3  121.03
#Mann= 3 , 0 , 0
   -12.9    .035       0       0    .035       0      11    .035       0
#XS Ineff= 2 , 0
               0  121.93      11          121.83
Permanent Ineff=
       F       F
Bank Sta=0,11
XS Rating Curve= 0
Exp/Cntr=.3,.1

Type RM Length L Ch R = 1 ,1409.00 ,16,16,16
BEGIN DESCRIPTION:
27.016
END DESCRIPTION:
#Sta/Elev= 21
    -9.1  119.06    -4.1  118.86    -4.1  119.66    -2.5  120.16       0  120.36
     1.4  120.16     1.4  119.76     2.9  119.76     2.9  119.16     3.4  119.16
     3.4  119.76     3.7  119.76     3.7  119.16     4.2  119.16     4.2  119.76
     6.1  119.76     6.6  119.36     7.1  119.36     7.6  119.76     8.5  119.76
    10.8  122.56
#Mann= 3 , 0 , 0
    -9.1    .035       0     1.4    .035       0     7.6    .035       0
#XS Ineff= 2 , 0
             1.4  120.16     7.6          119.76
Permanent Ineff=
       F       F
Bank Sta=1.4,7.6
XS Rating Curve= 0
Exp/Cntr=.3,.1

Type RM Length L Ch R = 1 ,1393.00 ,50,50,50
BEGIN DESCRIPTION:
27
END DESCRIPTION:
#Sta/Elev= 14
   -13.8  119.61    -3.8  119.61    -2.5  120.81       0  120.81     3.2  117.71
     7.4  117.71     8.2  119.81    10.2  120.81    12.7  120.81    13.5  119.81
    13.8  119.81      14  120.01    14.1  119.81    24.1  119.81
#Mann= 3 , 0 , 0
   -13.8    .035       0       0    .035       0    10.2    .035       0
#XS Ineff= 2 , 0
               0  120.81    10.2          120.81
Permanent Ineff=
       F       F
Bank Sta=0,10.2
XS Rating Curve= 0
Exp/Cntr=.3,.1

Type RM Length L Ch R = 1 ,1343.00 ,9,9,9
BEGIN DESCRIPTION:
26
END DESCRIPTION:
#Sta/Elev= 14
   -13.8  117.72    -3.8  117.72    -2.5  118.92       0  118.92     3.2  117.22
     7.4  117.22     8.2  117.92    10.2  118.92    12.7  118.92    13.5  117.92
    13.8  117.92      14  118.12    14.1  117.92    24.1  117.92
#Mann= 3 , 0 , 0
   -13.8    .035       0       0    .035       0    10.2    .035       0
#XS Ineff= 2 , 0
               0  118.92    10.2          118.92
Permanent Ineff=
       F       F
Bank Sta=0,10.2
XS Rating Curve= 0
Exp/Cntr=.3,.1

Type RM Length L Ch R = 1 ,1334.00 ,1,1,1
BEGIN DESCRIPTION:
25.041
END DESCRIPTION:
#Sta/Elev= 10
   -14.6  117.65    -4.6  117.65    -2.8  118.65       0  118.65     2.3  117.15
       7  117.15     9.1  118.65    11.4  118.35    13.1  117.75    23.1  117.75
#Mann= 3 , 0 , 0
   -14.6    .035       0       0    .035       0     9.1    .035       0
#XS Ineff= 2 , 0
               0  118.65     9.1          118.65
Permanent Ineff=
       F       F
Bank Sta=0,9.1
XS Rating Curve= 0
Exp/Cntr=.3,.1

Type RM Length L Ch R = 1 ,1333.00 ,22,22,22
BEGIN DESCRIPTION:
25.04
END DESCRIPTION:
#Sta/Elev= 12
   -14.6  117.65    -4.6  117.65    -2.8  118.65       0  118.65     2.3  117.15
     2.3  116.25       7  116.25       7  117.15     9.1  118.65    11.4  118.35
    13.1  117.75    23.1  117.75
#Mann= 3 , 0 , 0
   -14.6    .035       0       0    .035       0     9.1    .035       0
#XS Ineff= 2 , 0
               0  118.65     9.1          118.65
Permanent Ineff=
       F       F
Bank Sta=0,9.1
XS Rating Curve= 0
Exp/Cntr=.3,.1

Type RM Length L Ch R = 1 ,1311.00 ,18,18,18
BEGIN DESCRIPTION:
25.018
END DESCRIPTION:
#Sta/Elev= 14
   -15.2  116.29    -5.2  116.29    -3.2  117.79       0  117.79     2.8  115.99
     3.9  115.99     4.1  116.49     6.2  116.49     6.3  116.59     8.4  116.59
     9.5  117.59      12  117.59    12.5  117.19    22.5  117.19
#Mann= 3 , 0 , 0
   -15.2    .035       0       0    .035       0     9.5    .035       0
#XS Ineff= 2 , 0
               0  117.79     9.5          117.59
Permanent Ineff=
       F       F
Bank Sta=0,9.5
XS Rating Curve= 0
Exp/Cntr=.3,.1

Type RM Length L Ch R = 1 ,1293.00 ,2,2,2
BEGIN DESCRIPTION:
25
END DESCRIPTION:
#Sta/Elev= 9
    -4.3  116.31      -3  117.31       0  117.31     2.7  115.91     7.5  115.91
     8.9  117.21    11.9  117.21    12.6  116.51    22.6  116.51
#Mann= 3 , 0 , 0
    -4.3    .035       0       0    .035       0     8.9    .035       0
#XS Ineff= 2 , 0
               0  117.31     8.9          117.21
Permanent Ineff=
       F       F
Bank Sta=0,8.9
XS Rating Curve= 0
Exp/Cntr=.3,.1

Type RM Length L Ch R = 1 ,1291.00 ,10,10,10
BEGIN DESCRIPTION:
24.048
END DESCRIPTION:
#Sta/Elev= 9
    -4.3  116.25      -3  117.25       0  117.25     2.7  115.85     7.5  115.85
     8.9  117.15    11.9  117.15    12.6  116.45    22.6  116.45
#Mann= 3 , 0 , 0
    -4.3    .035       0       0    .035       0     8.9    .035       0
#XS Ineff= 2 , 0
               0  117.25     8.9          117.15
Permanent Ineff=
       F       F
Bank Sta=0,8.9
XS Rating Curve= 0
Exp/Cntr=.3,.1

Type RM Length L Ch R = 1 ,1281.00 ,38,38,38
BEGIN DESCRIPTION:
24.038
END DESCRIPTION:
#Sta/Elev= 8
     -10  116.84       0  116.84      .9  115.84     1.2  114.24    10.1  114.24
    10.4  115.94    11.7  116.84    21.7  116.84
#Mann= 3 , 0 , 0
     -10    .035       0       0    .035       0    11.7    .035       0
#XS Ineff= 2 , 0
               0  116.84    11.7          116.84
Permanent Ineff=
       F       F
Bank Sta=0,11.7
XS Rating Curve= 0
Exp/Cntr=.3,.1

Type RM Length L Ch R = 1 ,1243.00 ,12,12,12
BEGIN DESCRIPTION:
24
END DESCRIPTION:
#Sta/Elev= 12
   -12.8  114.76    -2.8  114.76    -1.8  115.56       0  115.56     2.1  114.16
     3.7  114.16     4.3  113.86     7.3  113.86    10.1  115.56    13.1  115.56
    13.5  115.16    23.5  115.16
#Mann= 3 , 0 , 0
   -12.8    .035       0       0    .035       0    10.1    .035       0
#XS Ineff= 2 , 0
               0  115.56    10.1          115.56
Permanent Ineff=
       F       F
Bank Sta=0,10.1
XS Rating Curve= 0
Exp/Cntr=.3,.1

Type RM Length L Ch R = 1 ,1231.00 ,1,1,1
BEGIN DESCRIPTION:
23.038
END DESCRIPTION:
#Sta/Elev= 14
   -13.6  114.85    -3.6  114.85      -2  115.35       0  115.35      .9  114.85
       3  113.65     6.2  113.65     6.4  114.05     6.6  114.55     8.7  114.55
      11  115.85    13.4  115.85    13.8  115.55    23.8  115.55
#Mann= 3 , 0 , 0
   -13.6    .035       0       0    .035       0      11    .035       0
#XS Ineff= 2 , 0
               0  115.35      11          115.85
Permanent Ineff=
       F       F
Bank Sta=0,11
XS Rating Curve= 0
Exp/Cntr=.3,.1

Type RM Length L Ch R = 1 ,1230.00 ,37,37,37
BEGIN DESCRIPTION:
23.037
END DESCRIPTION:
#Sta/Elev= 16
   -13.6  114.84    -3.6  114.85      -2  115.35       0  115.35      .9  114.85
       3  113.65       3  112.85     6.2  112.85     6.2  113.65     6.4  114.05
     6.6  114.55     8.7  114.55      11  115.85    13.4  115.85    13.8  115.55
    23.8  115.55
#Mann= 3 , 0 , 0
   -13.6    .035       0       0    .035       0      11    .035       0
#XS Ineff= 2 , 0
               0  115.35      11          115.85
Permanent Ineff=
       F       F
Bank Sta=0,11
XS Rating Curve= 0
Exp/Cntr=.3,.1

Type RM Length L Ch R = 1 ,1193.00 ,14,14,14
BEGIN DESCRIPTION:
23
END DESCRIPTION:
#Sta/Elev= 8
   -15.8  112.07    -5.8  112.07    -3.6  114.47       0  114.47     2.7  112.77
     7.7  112.77     8.7  114.37    18.7  114.37
#Mann= 3 , 0 , 0
   -15.8    .035       0       0    .035       0     8.7    .035       0
#XS Ineff= 2 , 0
               0  114.47     8.7          114.37
Permanent Ineff=
       F       F
Bank Sta=0,8.7
XS Rating Curve= 0
Exp/Cntr=.3,.1

Type RM Length L Ch R = 1 ,1179.00 ,36,36,36
BEGIN DESCRIPTION:
22.036
END DESCRIPTION:
#Sta/Elev= 8
   -15.8  111.83    -5.8  111.83    -3.6  114.23       0  114.23     2.7  112.53
     7.7  112.53     8.7  114.13    18.7  114.13
#Mann= 3 , 0 , 0
   -15.8    .035       0       0    .035       0     8.7    .035       0
#XS Ineff= 2 , 0
               0  114.23     8.7          114.13
Permanent Ineff=
       F       F
Bank Sta=0,8.7
XS Rating Curve= 0
Exp/Cntr=.3,.1

Type RM Length L Ch R = 1 ,1143.00 ,39,39,39
BEGIN DESCRIPTION:
22
END DESCRIPTION:
#Sta/Elev= 11
   -13.7  111.79    -3.7  111.79    -2.2  113.19       0  113.19     2.4  111.99
     3.7  111.69     7.7  111.69      10  112.89      13  112.89    13.3  112.59
    23.3  22.036
#Mann= 3 , 0 , 0
   -13.7    .035       0       0    .035       0      10    .035       0
#XS Ineff= 2 , 0
               0  113.19      10          112.89
Permanent Ineff=
       F       F
Bank Sta=0,10
XS Rating Curve= 0
Exp/Cntr=.3,.1

Type RM Length L Ch R = 1 ,1104.00 ,1,1,1
BEGIN DESCRIPTION:
21.011
END DESCRIPTION:
#Sta/Elev= 10
   -15.1  111.02    -5.1  111.02      -3  112.32       0  112.32     1.6  111.62
     9.6  111.62     9.6  112.02    12.6  112.02    12.9  111.92    22.9  111.92
#Mann= 3 , 0 , 0
   -15.1    .035       0       0    .035       0     9.6    .035       0
#XS Ineff= 2 , 0
               0  112.32     9.6          112.02
Permanent Ineff=
       F       F
Bank Sta=0,9.6
XS Rating Curve= 0
Exp/Cntr=.3,.1

Type RM Length L Ch R = 1 ,1103.00 ,10,10,10
BEGIN DESCRIPTION:
21.01
END DESCRIPTION:
#Sta/Elev= 12
   -15.1  111.02    -5.1  111.02      -3  112.32       0  112.32     1.6  111.62
     1.6  111.12     9.6  111.12     9.6  111.62     9.6  112.02    12.6  112.02
    12.9  111.92    22.9  111.92
#Mann= 3 , 0 , 0
   -15.1    .035       0       0    .035       0     9.6    .035       0
#XS Ineff= 2 , 0
               0  112.32     9.6          112.02
Permanent Ineff=
       F       F
Bank Sta=0,9.6
XS Rating Curve= 0
Exp/Cntr=.3,.1

Type RM Length L Ch R = 1 ,1093.00 ,39,39,39
BEGIN DESCRIPTION:
21
END DESCRIPTION:
#Sta/Elev= 11
   -12.9  111.47    -2.9  111.47    -2.3  111.87       0  111.87     2.1  111.07
     4.2  109.47       9  109.47    11.5  111.27    14.5  111.27    14.7  111.07
    24.7  111.07
#Mann= 3 , 0 , 0
   -12.9    .035       0       0    .035       0    11.5    .035       0
#XS Ineff= 2 , 0
               0  111.87    11.5          111.27
Permanent Ineff=
       F       F
Bank Sta=0,11.5
XS Rating Curve= 0
Exp/Cntr=.3,.1

Type RM Length L Ch R = 1 ,1054.00 ,11,11,11
BEGIN DESCRIPTION:
20.011
END DESCRIPTION:
#Sta/Elev= 11
   -12.9  110.25    -2.9  110.25    -2.3  110.65       0  110.65     2.1  110.25
     4.2  109.15       9  109.15    11.5  110.55    14.5  110.55    14.7  110.35
    24.7  110.35
#Mann= 3 , 0 , 0
   -12.9    .035       0       0    .035       0    11.5    .035       0
#XS Ineff= 2 , 0
               0  110.65    11.5          110.55
Permanent Ineff=
       F       F
Bank Sta=0,11.5
XS Rating Curve= 0
Exp/Cntr=.3,.1

Type RM Length L Ch R = 1 ,1043.00 ,50,50,50
BEGIN DESCRIPTION:
20
END DESCRIPTION:
#Sta/Elev= 14
   -13.4  109.23    -3.4  109.23    -2.2  110.33       0  110.33       3  108.13
     4.5  108.13     4.8  107.83     7.8  107.83     8.1  108.23     9.3  108.33
    11.9  110.23    14.3  110.23    14.5  110.03    24.5  110.03
#Mann= 3 , 0 , 0
   -13.4    .035       0       0    .035       0    11.9    .035       0
#XS Ineff= 2 , 0
               0  110.33    11.9          110.23
Permanent Ineff=
       F       F
Bank Sta=0,11.9
XS Rating Curve= 0
Exp/Cntr=.3,.1

Type RM Length L Ch R = 1 ,993.00  ,12,12,12
BEGIN DESCRIPTION:
19
END DESCRIPTION:
#Sta/Elev= 9
    -2.8  108.33    -2.5  108.63       0  108.63     2.2  106.93     6.8  106.93
     8.9  108.83    11.5  108.83    11.8  108.43    21.8  108.43
#Mann= 3 , 0 , 0
    -2.8    .035       0       0    .035       0     8.9    .035       0
#XS Ineff= 2 , 0
               0  108.63     8.9          108.83
Permanent Ineff=
       F       F
Bank Sta=0,8.9
XS Rating Curve= 0
Exp/Cntr=.3,.1

Type RM Length L Ch R = 1 ,981.00  ,28,28,28
BEGIN DESCRIPTION:
18.038
END DESCRIPTION:
#Sta/Elev= 9
    -2.8  108.02    -2.5  108.32       0  108.32     2.2  107.22     6.8  107.22
     8.9  108.52    11.5  108.52    11.8  108.12    21.8  108.12
#Mann= 3 , 0 , 0
    -2.8    .035       0       0    .035       0     8.9    .035       0
#XS Ineff= 2 , 0
               0  108.32     8.9          108.52
Permanent Ineff=
       F       F
Bank Sta=0,8.9
XS Rating Curve= 0
Exp/Cntr=.3,.1

Type RM Length L Ch R = 1 ,953.00  ,2,2,2
BEGIN DESCRIPTION:
18.01
END DESCRIPTION:
#Sta/Elev= 6
     -10  108.47       0  108.47     2.7  105.67    10.1  105.67    11.6  108.37
    21.6  108.37
#Mann= 3 , 0 , 0
     -10    .035       0       0    .035       0    11.6    .035       0
#XS Ineff= 2 , 0
               0  108.47    11.6          108.37
Permanent Ineff=
       F       F
Bank Sta=0,11.6
XS Rating Curve= 0
Exp/Cntr=.3,.1

Type RM Length L Ch R = 1 ,951.00  ,1,1,1
BEGIN DESCRIPTION:
18.008
END DESCRIPTION:
#Sta/Elev= 12
   -14.2  106.76    -9.2  106.86    -4.2  106.96    -4.2  108.16       0  108.16
      .7  107.46     2.6  105.56     7.5  105.56    10.2  107.16    12.9  107.16
    15.4  105.16    25.4  105.16
#Mann= 3 , 0 , 0
   -14.2    .035       0       0    .035       0    10.2    .035       0
#XS Ineff= 2 , 0
               0  108.16    10.2          107.16
Permanent Ineff=
       F       F
Bank Sta=0,10.2
XS Rating Curve= 0
Exp/Cntr=.3,.1

Type RM Length L Ch R = 1 ,950.00  ,50,50,50
BEGIN DESCRIPTION:
18.007
END DESCRIPTION:
#Sta/Elev= 13
    -9.2  106.86    -4.2  106.96    -4.2  108.16       0  108.16      .7  107.46
     2.6  105.56     2.6  105.06     7.5  105.06     7.5  105.56    10.2  107.16
    12.9  107.16    15.4  105.16    25.4  105.16
#Mann= 3 , 0 , 0
    -9.2    .035       0       0    .035       0    10.2    .035       0
#XS Ineff= 2 , 0
               0  108.16    10.2          107.16
Permanent Ineff=
       F       F
Bank Sta=0,10.2
XS Rating Curve= 0
Exp/Cntr=.3,.1

Type RM Length L Ch R = 1 ,900.00  ,50,50,50
BEGIN DESCRIPTION:
18
END DESCRIPTION:
#Sta/Elev= 14
   -16.5  106.18    -6.5  106.18    -6.1  106.78    -4.6  106.78    -2.2  107.88
       0  107.88     2.7  105.68     4.4  105.38     5.4  105.38     8.2  105.88
     9.9  107.28    12.9  107.28    14.2  105.68    24.2  105.68
#Mann= 3 , 0 , 0
   -16.5    .035       0       0    .035       0     9.9    .035       0
#XS Ineff= 2 , 0
               0  107.88     9.9          107.28
Permanent Ineff=
       F       F
Bank Sta=0,9.9
XS Rating Curve= 0
Exp/Cntr=.3,.1

Type RM Length L Ch R = 1 ,850.00  ,50,50,50
BEGIN DESCRIPTION:
17
END DESCRIPTION:
#Sta/Elev= 12
   -13.1  105.83    -3.1  105.83    -2.5  106.23       0  106.23     3.5  104.83
       9  104.83     9.5  104.63    10.5  104.63      13  106.63    15.5  106.63
    16.2  106.03    26.2  106.03
#Mann= 3 , 0 , 0
   -13.1    .035       0       0    .035       0      13    .035       0
#XS Ineff= 2 , 0
               0  106.23      13          106.63
Permanent Ineff=
       F       F
Bank Sta=0,13
XS Rating Curve= 0
Exp/Cntr=.3,.1

Type RM Length L Ch R = 1 ,800.00  ,10,10,10
BEGIN DESCRIPTION:
16
END DESCRIPTION:
#Sta/Elev= 12
   -13.1  105.83    -3.1  105.83    -2.5  106.23       0  106.23     3.5  104.83
       9  104.83     9.5  104.63    10.5  104.63      13  106.63    15.5  106.63
    16.2  106.03    26.2  106.03
#Mann= 3 , 0 , 0
   -13.1    .035       0       0    .035       0      13    .035       0
#XS Ineff= 2 , 0
               0  106.23      13          106.63
Permanent Ineff=
       F       F
Bank Sta=0,13
XS Rating Curve= 0
Exp/Cntr=.3,.1

Type RM Length L Ch R = 1 ,790.00  ,1,1,1
BEGIN DESCRIPTION:
15.04
END DESCRIPTION:
#Sta/Elev= 9
   -12.9  105.17    -2.9  105.17    -2.5  105.47       0  105.47     1.8  104.47
     3.8  103.67     9.6  103.67    12.9  104.87    22.9  104.87
#Mann= 3 , 0 , 0
   -12.9    .035       0       0    .035       0    12.9    .035       0
#XS Ineff= 2 , 0
               0  105.47    12.9          104.87
Permanent Ineff=
       F       F
Bank Sta=0,12.9
XS Rating Curve= 0
Exp/Cntr=.3,.1

Type RM Length L Ch R = 1 ,789.00  ,15,15,15
BEGIN DESCRIPTION:
15.039
END DESCRIPTION:
#Sta/Elev= 11
   -12.9  105.17    -2.9  105.17    -2.5  105.47       0  105.47     1.8  104.47
     3.8  103.67     3.8  102.17     9.6  102.17     9.6  103.67    12.9  104.87
    22.9  104.87
#Mann= 3 , 0 , 0
   -12.9    .035       0       0    .035       0    12.9    .035       0
#XS Ineff= 2 , 0
               0  105.47    12.9          104.87
Permanent Ineff=
       F       F
Bank Sta=0,12.9
XS Rating Curve= 0
Exp/Cntr=.3,.1

Type RM Length L Ch R = 1 ,774.00  ,24,24,24
BEGIN DESCRIPTION:
15.024
END DESCRIPTION:
#Sta/Elev= 11
     -10  105.37       0  105.37     4.7  102.67     6.5  102.67       8  101.97
     9.5  101.97    11.2  102.87    14.6  105.57    17.7  105.57    20.2  104.37
    30.2  104.37
#Mann= 3 , 0 , 0
     -10    .035       0       0    .035       0    14.6    .035       0
#XS Ineff= 2 , 0
               0  105.37    14.6          105.57
Permanent Ineff=
       F       F
Bank Sta=0,14.6
XS Rating Curve= 0
Exp/Cntr=.3,.1

Type RM Length L Ch R = 1 ,750.00  ,50,50,50
BEGIN DESCRIPTION:
15
END DESCRIPTION:
#Sta/Elev= 10
   -12.5  104.54    -2.5  104.54      -2  104.94       0  104.94     3.2  101.74
    10.2  101.74    13.4  104.94    16.1  104.94    16.5  104.64    26.5  104.64
#Mann= 3 , 0 , 0
   -12.5    .035       0       0    .035       0    13.4    .035       0
#XS Ineff= 2 , 0
               0  104.94    13.4          104.94
Permanent Ineff=
       F       F
Bank Sta=0,13.4
XS Rating Curve= 0
Exp/Cntr=.3,.1

Type RM Length L Ch R = 1 ,700.00  ,30,30,30
BEGIN DESCRIPTION:
14
END DESCRIPTION:
#Sta/Elev= 10
   -12.5  103.65    -2.5  103.65      -2  104.05       0  104.05     3.2  101.25
    10.2  101.25    13.4  104.05    16.1  104.05    16.5  103.75    26.5  103.75
#Mann= 3 , 0 , 0
   -12.5    .035       0       0    .035       0    13.4    .035       0
#XS Ineff= 2 , 0
               0  104.05    13.4          104.05
Permanent Ineff=
       F       F
Bank Sta=0,13.4
XS Rating Curve= 0
Exp/Cntr=.3,.1

Type RM Length L Ch R = 1 ,670.00  ,20,20,20
BEGIN DESCRIPTION:
13.02
END DESCRIPTION:
#Sta/Elev= 9
     -10  103.64       0  103.64     2.5  101.34     7.7  101.34    10.7  103.94
    13.9  106.34    16.6  106.34    18.2  104.64    28.2  104.64
#Mann= 3 , 0 , 0
     -10    .035       0       0    .035       0    13.9    .035       0
#XS Ineff= 2 , 0
               0  103.64    13.9          106.34
Permanent Ineff=
       F       F
Bank Sta=0,13.9
XS Rating Curve= 0
Exp/Cntr=.3,.1

Type RM Length L Ch R = 1 ,650.00  ,50,50,50
BEGIN DESCRIPTION:
13
END DESCRIPTION:
#Sta/Elev= 12
   -11.9  102.74    -1.9  102.74    -1.5  103.04       0  103.04     3.4  100.84
       6  100.24     9.7  100.24    10.7  100.64    14.1  102.54    17.1  102.54
    17.5  102.24    27.5  102.24
#Mann= 3 , 0 , 0
   -11.9    .035       0       0    .035       0    14.1    .035       0
#XS Ineff= 2 , 0
               0  103.04    14.1          102.54
Permanent Ineff=
       F       F
Bank Sta=0,14.1
XS Rating Curve= 0
Exp/Cntr=.3,.1

Type RM Length L Ch R = 1 ,600.00  ,22,22,22
BEGIN DESCRIPTION:
12
END DESCRIPTION:
#Sta/Elev= 12
   -11.9  102.38    -1.9  102.38    -1.5  102.68       0  102.68     3.4  100.38
       6   99.78     9.7   99.78    10.7  100.18    14.1  102.18    17.1  102.18
    17.5  101.88    27.5  101.88
#Mann= 3 , 0 , 0
   -11.9    .035       0       0    .035       0    14.1    .035       0
#XS Ineff= 2 , 0
               0  102.68    14.1          102.18
Permanent Ineff=
       F       F
Bank Sta=0,14.1
XS Rating Curve= 0
Exp/Cntr=.3,.1

Type RM Length L Ch R = 1 ,578.00  ,28,28,28
BEGIN DESCRIPTION:
11.028
END DESCRIPTION:
#Sta/Elev= 8
     -10  102.62       0  102.62     2.5  100.22     4.7   99.82     7.7   99.82
      10  100.12    12.7  102.82    22.7  102.82
#Mann= 3 , 0 , 0
     -10    .035       0       0    .035       0    12.7    .035       0
#XS Ineff= 2 , 0
               0  102.62    12.7          102.82
Permanent Ineff=
       F       F
Bank Sta=0,12.7
XS Rating Curve= 0
Exp/Cntr=.3,.1

Type RM Length L Ch R = 1 ,550.00  ,50,50,50
BEGIN DESCRIPTION:
11
END DESCRIPTION:
#Sta/Elev= 13
   -13.4  101.19    -3.4  101.19    -2.6  102.09       0  102.09       3  100.29
     5.3   99.89     5.9   99.49     8.6   99.49    11.1  101.19    12.6  101.49
    14.9  101.49    15.5  100.99    25.5  100.99
#Mann= 3 , 0 , 0
   -13.4    .035       0       0    .035       0    12.6    .035       0
#XS Ineff= 2 , 0
               0  102.09    12.6          101.49
Permanent Ineff=
       F       F
Bank Sta=0,12.6
XS Rating Curve= 0
Exp/Cntr=.3,.1

Type RM Length L Ch R = 1 ,500.00  ,18,18,18
BEGIN DESCRIPTION:
10
END DESCRIPTION:
#Sta/Elev= 13
   -13.4  100.26    -3.4  100.26    -2.6  101.16       0  101.16       3   99.56
     5.3   99.36     5.9   99.06     8.6   99.06    11.1  100.66    12.6  100.96
    14.9  100.96    15.5  100.46    25.5  100.46
#Mann= 3 , 0 , 0
   -13.4    .035       0       0    .035       0    12.6    .035       0
#XS Ineff= 2 , 0
               0  101.16    12.6          100.96
Permanent Ineff=
       F       F
Bank Sta=0,12.6
XS Rating Curve= 0
Exp/Cntr=.3,.1

Type RM Length L Ch R = 1 ,482.00  ,32,32,32
BEGIN DESCRIPTION:
9.032
END DESCRIPTION:
#Sta/Elev= 10
   -12.9  100.48    -2.9  100.48    -2.5  100.78       0  100.78     2.3   97.88
     8.3   97.88    11.8   99.38    14.4   99.38    14.9   99.08    24.9   99.08
#Mann= 3 , 0 , 0
   -12.9    .035       0       0    .035       0    11.8    .035       0
#XS Ineff= 2 , 0
               0  100.78    11.8           99.38
Permanent Ineff=
       F       F
Bank Sta=0,11.8
XS Rating Curve= 0
Exp/Cntr=.3,.1

Type RM Length L Ch R = 1 ,450.00  ,50,50,50
BEGIN DESCRIPTION:
9
END DESCRIPTION:
#Sta/Elev= 15
     -13   99.59      -3   99.59    -2.5  100.09       0  100.09     3.5   98.19
     5.7   97.79     6.1   97.29     9.1   97.29    10.6   97.99    13.6   98.49
    16.6  100.19    17.6  100.89    20.2  100.89    20.9  100.39    30.9  100.39
#Mann= 3 , 0 , 0
     -13    .035       0       0    .035       0    17.6    .035       0
#XS Ineff= 2 , 0
               0  100.09    17.6          100.89
Permanent Ineff=
       F       F
Bank Sta=0,17.6
XS Rating Curve= 0
Exp/Cntr=.3,.1

Type RM Length L Ch R = 1 ,400.00  ,50,50,50
BEGIN DESCRIPTION:
8
END DESCRIPTION:
#Sta/Elev= 14
     -13    99.2      -3    99.2    -2.5    99.7       0    99.7     3.5    97.8
     5.7    97.4     6.1    96.9     9.1    96.9    10.6    97.6    12.9    98.1
    15.9    98.8    18.5    98.8    19.2    98.3    29.2    98.3
#Mann= 3 , 0 , 0
     -13    .035       0       0    .035       0    15.9    .035       0
#XS Ineff= 2 , 0
               0    99.7    15.9            98.8
Permanent Ineff=
       F       F
Bank Sta=0,15.9
XS Rating Curve= 0
Exp/Cntr=.3,.1

Type RM Length L Ch R = 1 ,350.00  ,50,50,50
BEGIN DESCRIPTION:
7
END DESCRIPTION:
#Sta/Elev= 8
     -10   99.44       0   99.44     2.6   97.14     4.3   97.04     4.9   96.54
    11.8   96.54      15   98.64      25   98.64
#Mann= 3 , 0 , 0
     -10    .035       0       0    .035       0      15    .035       0
#XS Ineff= 2 , 0
               0   99.44      15           98.64
Permanent Ineff=
       F       F
Bank Sta=0,15
XS Rating Curve= 0
Exp/Cntr=.3,.1

Type RM Length L Ch R = 1 ,300.00  ,34,34,34
BEGIN DESCRIPTION:
6
END DESCRIPTION:
#Sta/Elev= 8
     -10   98.56       0   98.56     2.6   96.16     4.3   95.96     4.9   95.46
    11.8   95.46      15   97.66      25   97.66
#Mann= 3 , 0 , 0
     -10    .035       0       0    .035       0      15    .035       0
#XS Ineff= 2 , 0
               0   98.56      15           97.66
Permanent Ineff=
       F       F
Bank Sta=0,15
XS Rating Curve= 0
Exp/Cntr=.3,.1

Type RM Length L Ch R = 1 ,266.00  ,16,16,16
BEGIN DESCRIPTION:
5.016
END DESCRIPTION:
#Sta/Elev= 8
     -10    98.1       0    98.1     2.6    95.8     4.3    95.6     4.9    95.1
    11.8    95.1      15    97.2      25    97.2
#Mann= 3 , 0 , 0
     -10    .035       0       0    .035       0      15    .035       0
#XS Ineff= 2 , 0
               0    98.1      15            97.2
Permanent Ineff=
       F       F
Bank Sta=0,15
XS Rating Curve= 0
Exp/Cntr=.3,.1

Type RM Length L Ch R = 1 ,250.00  ,50,50,50
BEGIN DESCRIPTION:
5
END DESCRIPTION:
#Sta/Elev= 12
   -14.6    96.7    -4.6    96.7    -3.6      98       0      98     1.3    97.1
     4.3      95     9.8      95    12.8    97.1      14    97.9      17    97.9
    18.2    96.6    28.2    96.6
#Mann= 3 , 0 , 0
   -14.6    .035       0       0    .035       0      14    .035       0
#XS Ineff= 2 , 0
               0      98      14            97.9
Permanent Ineff=
       F       F
Bank Sta=0,14
XS Rating Curve= 0
Exp/Cntr=.3,.1

Type RM Length L Ch R = 1 ,200.00  ,50,50,50
BEGIN DESCRIPTION:
4
END DESCRIPTION:
#Sta/Elev= 12
   -13.6   96.96    -3.6   96.96    -2.9   97.56       0   97.56     2.7   94.66
     5.7   94.66     6.8   94.96    11.8   94.96    14.1   96.76    16.8   96.76
    17.8   95.86    27.8   95.86
#Mann= 3 , 0 , 0
   -13.6    .035       0       0    .035       0    14.1    .035       0
#XS Ineff= 2 , 0
               0   97.56    14.1           96.76
Permanent Ineff=
       F       F
Bank Sta=0,14.1
XS Rating Curve= 0
Exp/Cntr=.3,.1

Type RM Length L Ch R = 1 ,150.00  ,14,14,14
BEGIN DESCRIPTION:
3
END DESCRIPTION:
#Sta/Elev= 15
   -12.8      97    -2.8      97    -2.5    97.2       0    97.2       3    96.2
     4.5    95.1     5.8    95.1     6.1    94.5    10.4    94.5    11.1    95.2
    12.8    95.4    15.8    96.4    18.8    96.4    18.9    96.3    28.9    96.3
#Mann= 3 , 0 , 0
   -12.8    .035       0       0    .035       0    15.8    .035       0
#XS Ineff= 2 , 0
               0    97.2    15.8            96.4
Permanent Ineff=
       F       F
Bank Sta=0,15.8
XS Rating Curve= 0
Exp/Cntr=.3,.1

Type RM Length L Ch R = 1 ,136.00  ,36,36,36
BEGIN DESCRIPTION:
2.036
END DESCRIPTION:
#Sta/Elev= 15
   -12.8   96.92    -2.8   96.92    -2.5   97.12       0   97.12       3   96.12
     4.5   95.52     5.8   95.52     6.1   95.12    10.4   95.12    11.1   95.62
    12.8   95.82    15.8   97.52    18.8   97.52    18.9   97.42    28.9   97.42
#Mann= 3 , 0 , 0
   -12.8    .035       0       0    .035       0    15.8    .035       0
#XS Ineff= 2 , 0
               0   97.12    15.8           97.52
Permanent Ineff=
       F       F
Bank Sta=0,15.8
XS Rating Curve= 0
Exp/Cntr=.3,.1

Type RM Length L Ch R = 1 ,100.00  ,50,50,50
BEGIN DESCRIPTION:
2
END DESCRIPTION:
#Sta/Elev= 15
   -12.8   96.75    -2.8   96.75    -2.5   96.95       0   96.95       3   95.35
     4.5   94.35     5.8   94.35     6.1   93.85    10.4   93.85    11.1   94.45
    12.8   94.65    15.8   96.35    18.8   96.35    18.9   96.25    28.9   96.25
#Mann= 3 , 0 , 0
   -12.8    .035       0       0    .035       0    15.8    .035       0
#XS Ineff= 2 , 0
               0   96.95    15.8           96.35
Permanent Ineff=
       F       F
Bank Sta=0,15.8
XS Rating Curve= 0
Exp/Cntr=.3,.1

Type RM Length L Ch R = 1 ,50.00   ,13,13,13
BEGIN DESCRIPTION:
1
END DESCRIPTION:
#Sta/Elev= 6
     -10   96.58       0   96.58       0   93.48       9   93.48       9   96.58
      19   96.58
#Mann= 3 , 0 , 0
     -10    .035       0       0    .035       0       9    .035       0
#XS Ineff= 2 , 0
               0   96.58       9           96.58
Permanent Ineff=
       F       F
Bank Sta=0,9
XS Rating Curve= 0
Exp/Cntr=.3,.1

Type RM Length L Ch R = 1 ,37.00   ,21,21,21
BEGIN DESCRIPTION:
0.037
END DESCRIPTION:
#Sta/Elev= 6
     -10   96.44       0   96.44       0   93.24       9   93.24       9   96.44
      19   96.44
#Mann= 3 , 0 , 0
     -10    .035       0       0    .035       0       9    .035       0
#XS Ineff= 2 , 0
               0   96.44       9           96.44
Permanent Ineff=
       F       F
Bank Sta=0,9
XS Rating Curve= 0
Exp/Cntr=.3,.1

Type RM Length L Ch R = 1 ,16.00   ,16,16,16
BEGIN DESCRIPTION:
0.016
END DESCRIPTION:
#Sta/Elev= 6
     -10   96.64       0   96.64       0   93.04     7.8   93.04     7.8   96.44
    17.8   96.44
#Mann= 3 , 0 , 0
     -10    .035       0       0    .035       0     7.8    .035       0
#XS Ineff= 2 , 0
               0   96.64     7.8           96.44
Permanent Ineff=
       F       F
Bank Sta=0,7.8
XS Rating Curve= 0
Exp/Cntr=.3,.1

Type RM Length L Ch R = 1 ,0.00    ,0,0,0
BEGIN DESCRIPTION:
0
END DESCRIPTION:
#Sta/Elev= 12
     -10   96.42       0   96.42       3   94.32     4.1   94.32     7.1   93.12
     8.6   92.42    13.1   92.42    13.4   92.82    15.7   93.82    18.5   95.02
    21.6   96.32    31.6   96.32
#Mann= 3 , 0 , 0
     -10    .035       0       0    .035       0    21.6    .035       0
#XS Ineff= 2 , 0
               0   96.42    21.6           96.32
Permanent Ineff=
       F       F
Bank Sta=0,21.6
XS Rating Curve= 0
Exp/Cntr=.3,.1

Chan Stop Cuts=-1
