--- OKMA.prj (project) ---

Proj Title=OKMA
Current Plan=p01
Default Exp/Contr=.3,.1
SI Units
Geom File=g01
Flow File=f01
Plan File=p01
Y Axis Title=Elevation
X Axis Title(PF)=Main Channel Distance
X Axis Title(XS)=Station
BEGIN DESCRIPTION:
           BACK WATER COMPUTATION
      APPLICATION OF HEC-2 BY Samju Construction Engineering
      OKMA-STREEM : 30 YR
END DESCRIPTION:
DSS Export Rating Curves= 0
DSS Export Rating Curve Sorted= 0
DSS Export Volume Flow Curves= 0
DXF OffsetX= 0
DXF OffsetY= 0
DXF ScaleX= 1
DXF ScaleY= 10

--- OKMA.p01 (plan) ---

Plan Title=Imported Plan 01
Version=Version 3.0.1  Mar 2001
Short Identifier=Imported Pla
Geom File=g01
Flow File=f01
Subcritical Flow
K Sum by GR= 0
Std Step Tol= 0.003
Critical Tol= 0.003
Num of Std Step Trials= 20
Max Error Tol= 0.1
Flow Tol Ratio= 0.001
Split Flow NTrial= 30
Split Flow Tol= 0.02
Split Flow Ratio= 0.02
Log Output Level= 0
Friction Slope Method= 1
Unsteady Friction Slope Method= 2
Parabolic Critical Depth
Global Vel Dist= 0 , 0 , 0
Global Log Level= 0
CheckData=True
Encroach Param=-1 ,0,0, 0
Computation Interval=1HOUR
Output Interval=1HOUR
Run HTab= 0
Run UNet= 0
Run PostProcess= 0
UNET Theta= 1
UNET ZTol= 0.02
UNET ZSATol= 0.1
UNET MxIter= 20
UNET MaxInSteps= 20
UNET DtIC= 0
UNET DtMin= 0
UNET MaxCRTS= 20
UNET WFStab= 2
UNET SFStab= 1
UNET WFX= 1
UNET SFX= 1
UNET Convert EG Bridges=-1
UNET Use Existing IB Tables=-1
Instantaneous Interval=1HOUR
Write IC File= 0
Write Velocity= 0
Write Detailed= 0

--- OKMA.f01 (steady flow) ---

Flow Title=Imported Flow 01
Version=Version 3.0.1  Mar 2001
Number of Profiles= 5
Profile Names=10YR,20YR,30YR,50YR,80YR
River Rch & RM=RIVER-1,Reach-1         ,58.027
   16.24    17.9   18.87   20.09   21.21
River Rch & RM=RIVER-1,Reach-1         ,16.026
   18.87    20.8   21.93   23.36   24.67
River Rch & RM=OKMA,OKMA            ,2927.00
   16.24    17.9   18.87   20.09   21.21
River Rch & RM=OKMA,OKMA            ,826.00
   18.87    20.8   21.93   23.36   24.67
Boundary for River Rch & Prof#=OKMA,OKMA            , 1
Up Type= 0
Dn Type= 3
Dn Slope=.022
Boundary for River Rch & Prof#=OKMA,OKMA            , 2
Up Type= 0
Dn Type= 3
Dn Slope=.022
Boundary for River Rch & Prof#=OKMA,OKMA            , 3
Up Type= 0
Dn Type= 3
Dn Slope=.022
Boundary for River Rch & Prof#=OKMA,OKMA            , 4
Up Type= 0
Dn Type= 3
Dn Slope=.022
Boundary for River Rch & Prof#=OKMA,OKMA            , 5
Up Type= 0
Dn Type= 3
Dn Slope=.022
DSS Import GetInterval= 0
DSS Import GetPeak= 0
DSS Import FillOption= 0

--- OKMA.g01 (geometry) ---

Geom Title=Imported Geom 01
Version=Version 3.0.1  Mar 2001

River Reach=OKMA            ,OKMA
Reach XY= 2
              .5             .95              .5             .05

Type RM Length L Ch R = 1 ,2927.00 ,27,27,27
BEGIN DESCRIPTION:
58.027
END DESCRIPTION:
#Sta/Elev= 17
   -10.7   72.29     -.7   72.29     -.5   72.49       0   72.49     1.5   71.69
     1.9   71.69     2.6   72.09     2.8   72.09       4   71.39     4.7   70.39
     5.2   69.99     6.7   69.99     7.1   70.89     8.7   71.89    10.9   71.89
    12.4   70.69    22.4   70.69
#Mann= 3 , 0 , 0
   -10.7    .033       0       0    .033       0     8.7    .033       0
#XS Ineff= 2 , 0
               0   72.49     8.7           71.89
Permanent Ineff=
       F       F
Bank Sta=0,8.7
XS Rating Curve= 0
Exp/Cntr=.3,.1

Type RM Length L Ch R = 1 ,2900.00 ,30,30,30
BEGIN DESCRIPTION:
58
END DESCRIPTION:
#Sta/Elev= 8
     -10   70.25       0   70.25     1.3   69.25     1.8   68.65     2.2   68.65
     3.9   69.15     5.6   70.35    15.6   70.35
#Mann= 3 , 0 , 0
     -10    .033       0       0    .033       0     5.6    .033       0
#XS Ineff= 2 , 0
               0   70.25     5.6           70.35
Permanent Ineff=
       F       F
Bank Sta=0,5.6
XS Rating Curve= 0
Exp/Cntr=.3,.1

Type RM Length L Ch R = 1 ,2870.00 ,20,20,20
BEGIN DESCRIPTION:
57.02
END DESCRIPTION:
#Sta/Elev= 6
     -10   68.38       0   68.38      .1   67.28     2.5   67.28     2.6   68.38
    12.6   68.38
#Mann= 3 , 0 , 0
     -10    .033       0       0    .033       0     2.6    .033       0
#XS Ineff= 2 , 0
               0   68.38     2.6           68.38
Permanent Ineff=
       F       F
Bank Sta=0,2.6
XS Rating Curve= 0
Exp/Cntr=.3,.1

Type RM Length L Ch R = 1 ,2850.00 ,50,50,50
BEGIN DESCRIPTION:
57
END DESCRIPTION:
#Sta/Elev= 7
     -10   67.54       0   67.54      .2   66.44     2.1   66.44     2.5   67.64
     2.9   68.04    12.9   68.04
#Mann= 3 , 0 , 0
     -10    .033       0       0    .033       0     2.9    .033       0
#XS Ineff= 2 , 0
               0   67.54     2.9           68.04
Permanent Ineff=
       F       F
Bank Sta=0,2.9
XS Rating Curve= 0
Exp/Cntr=.3,.1

Type RM Length L Ch R = 1 ,2800.00 ,50,50,50
BEGIN DESCRIPTION:
56
END DESCRIPTION:
#Sta/Elev= 7
     -10   65.45       0   65.45      .2   64.25     2.1   64.25     2.5   65.45
     2.9   65.85    12.9   65.85
#Mann= 3 , 0 , 0
     -10    .033       0       0    .033       0     2.9    .033       0
#XS Ineff= 2 , 0
               0   65.45     2.9           65.85
Permanent Ineff=
       F       F
Bank Sta=0,2.9
XS Rating Curve= 0
Exp/Cntr=.3,.1

Type RM Length L Ch R = 1 ,2750.00 ,50,50,50
BEGIN DESCRIPTION:
55
END DESCRIPTION:
#Sta/Elev= 10
   -14.3   60.93    -4.3   60.93    -2.3   62.43      -1   62.43     -.6   62.23
       0   62.23      .3   61.43     3.3   61.43     3.3   63.03    13.3   63.03
#Mann= 3 , 0 , 0
   -14.3    .033       0       0    .033       0     3.3    .033       0
#XS Ineff= 2 , 0
               0   62.23     3.3           63.03
Permanent Ineff=
       F       F
Bank Sta=0,3.3
XS Rating Curve= 0
Exp/Cntr=.3,.1

Type RM Length L Ch R = 1 ,2700.00 ,50,50,50
BEGIN DESCRIPTION:
54
END DESCRIPTION:
#Sta/Elev= 10
   -14.3   58.98    -4.3   58.98    -2.3   60.48      -1   60.48     -.6   60.28
       0   60.28      .3   59.38     3.3   59.38     3.3   60.98    13.3   60.98
#Mann= 3 , 0 , 0
   -14.3    .033       0       0    .033       0     3.3    .033       0
#XS Ineff= 2 , 0
               0   60.28     3.3           60.98
Permanent Ineff=
       F       F
Bank Sta=0,3.3
XS Rating Curve= 0
Exp/Cntr=.3,.1

Type RM Length L Ch R = 1 ,2650.00 ,50,50,50
BEGIN DESCRIPTION:
53
END DESCRIPTION:
#Sta/Elev= 10
   -14.3   57.31    -4.3   57.31    -2.3   58.81      -1   58.81     -.6   58.61
       0   58.61      .3   57.01     3.3   57.01     3.3   59.11    13.3   59.11
#Mann= 3 , 0 , 0
   -14.3    .033       0       0    .033       0     3.3    .033       0
#XS Ineff= 2 , 0
               0   58.61     3.3           59.11
Permanent Ineff=
       F       F
Bank Sta=0,3.3
XS Rating Curve= 0
Exp/Cntr=.3,.1

Type RM Length L Ch R = 1 ,2600.00 ,50,50,50
BEGIN DESCRIPTION:
52
END DESCRIPTION:
#Sta/Elev= 8
   -14.5   56.17    -4.5   56.17    -3.5   57.37       0   57.37      .3   55.77
     2.5    55.7       3   58.07      13   58.07
#Mann= 3 , 0 , 0
   -14.5    .033       0       0    .033       0       3    .033       0
#XS Ineff= 2 , 0
               0   57.37       3           58.07
Permanent Ineff=
       F       F
Bank Sta=0,3
XS Rating Curve= 0
Exp/Cntr=.3,.1

Type RM Length L Ch R = 1 ,2550.00 ,10,10,10
BEGIN DESCRIPTION:
51
END DESCRIPTION:
#Sta/Elev= 8
   -14.5   54.53    -4.5   54.53      -3   55.73       0   55.73      .3   54.43
     2.5   54.43       3   56.43      13   56.43
#Mann= 3 , 0 , 0
   -14.5    .033       0       0    .033       0       3    .033       0
#XS Ineff= 2 , 0
               0   55.73       3           56.43
Permanent Ineff=
       F       F
Bank Sta=0,3
XS Rating Curve= 0
Exp/Cntr=.3,.1

Type RM Length L Ch R = 1 ,2540.00 ,40,40,40
BEGIN DESCRIPTION:
50.04
END DESCRIPTION:
#Sta/Elev= 9
   -14.5   54.43    -4.5   54.43      -3   55.43       0   55.43      .5   54.33
     1.2   54.23     2.5   54.23       3   55.63      13   55.63
#Mann= 3 , 0 , 0
   -14.5    .033       0       0    .033       0       3    .033       0
#XS Ineff= 2 , 0
               0   55.43       3           55.63
Permanent Ineff=
       F       F
Bank Sta=0,3
XS Rating Curve= 0
Exp/Cntr=.3,.1

Type RM Length L Ch R = 1 ,2500.00 ,27,27,27
BEGIN DESCRIPTION:
50
END DESCRIPTION:
#Sta/Elev= 11
   -15.2   51.61    -5.2   51.61      -5   52.71      -3   54.21       0   54.21
      .4   53.21     1.2   53.21     1.4   53.71     2.2   53.71     2.6   54.41
    12.6   54.41
#Mann= 3 , 0 , 0
   -15.2    .033       0       0    .033       0     2.6    .033       0
#XS Ineff= 2 , 0
               0   54.21     2.6           54.41
Permanent Ineff=
       F       F
Bank Sta=0,2.6
XS Rating Curve= 0
Exp/Cntr=.3,.1

Type RM Length L Ch R = 1 ,2473.00 ,23,23,23
BEGIN DESCRIPTION:
49.023
END DESCRIPTION:
#Sta/Elev= 8
     -14   52.54      -4   52.54    -2.8   53.54       0   53.84      .3   52.44
     2.2   52.44     2.6   53.74    12.6   53.74
#Mann= 3 , 0 , 0
     -14    .033       0       0    .033       0     2.6    .033       0
#XS Ineff= 2 , 0
               0   53.84     2.6           53.74
Permanent Ineff=
       F       F
Bank Sta=0,2.6
XS Rating Curve= 0
Exp/Cntr=.3,.1

Type RM Length L Ch R = 1 ,2450.00 ,50,50,50
BEGIN DESCRIPTION:
49
END DESCRIPTION:
#Sta/Elev= 14
   -13.2   51.19    -3.2   51.19    -1.6   52.39     -.6   52.59     -.6   52.69
       0   52.69      .4   51.29     1.4   51.29     1.5   51.89     2.6   51.99
     2.9   52.79     5.5   52.79     7.1   51.79    17.1   51.79
#Mann= 3 , 0 , 0
   -13.2    .033       0       0    .033       0     2.9    .033       0
#XS Ineff= 2 , 0
               0   52.69     2.9           52.79
Permanent Ineff=
       F       F
Bank Sta=0,2.9
XS Rating Curve= 0
Exp/Cntr=.3,.1

Type RM Length L Ch R = 1 ,2400.00 ,39,39,39
BEGIN DESCRIPTION:
48
END DESCRIPTION:
#Sta/Elev= 14
     -10   49.91    -3.2   49.91    -1.6   51.11     -.6   51.31     -.6   51.41
       0   51.41      .4   50.01     1.4   50.01     1.5   50.61     2.6   50.71
     2.9   51.51     5.5   51.51     7.1   50.51    17.1   50.51
#Mann= 3 , 0 , 0
     -10    .033       0       0    .033       0     2.9    .033       0
#XS Ineff= 2 , 0
               0   51.41     2.9           51.51
Permanent Ineff=
       F       F
Bank Sta=0,2.9
XS Rating Curve= 0
Exp/Cntr=.3,.1

Type RM Length L Ch R = 1 ,2361.00 ,11,11,11
BEGIN DESCRIPTION:
47.011
END DESCRIPTION:
#Sta/Elev= 14
   -13.8   48.68    -3.8   48.68      -2   50.28       0   50.28      .2   49.08
      .5   49.08      .5   48.88     1.9   48.88     1.9   49.08     2.1   49.08
     2.5   50.28       5   50.28     6.2   49.18    16.2   49.18
#Mann= 3 , 0 , 0
   -13.8    .033       0       0    .033       0     2.5    .033       0
#XS Ineff= 2 , 0
               0   50.28     2.5           50.28
Permanent Ineff=
       F       F
Bank Sta=0,2.5
XS Rating Curve= 0
Exp/Cntr=.3,.1

Type RM Length L Ch R = 1 ,2350.00 ,50,50,50
BEGIN DESCRIPTION:
47
END DESCRIPTION:
#Sta/Elev= 14
   -12.2   48.29    -3.8   48.29      -2   49.89       0   49.89      .2   48.69
      .5   48.69      .5   48.49     1.9   48.49     1.9   48.69     2.1   48.69
     2.5   49.89       5   49.89     6.2   48.79    16.2   48.79
#Mann= 3 , 0 , 0
   -12.2    .033       0       0    .033       0     2.5    .033       0
#XS Ineff= 2 , 0
               0   49.89     2.5           49.89
Permanent Ineff=
       F       F
Bank Sta=0,2.5
XS Rating Curve= 0
Exp/Cntr=.3,.1

Type RM Length L Ch R = 1 ,2300.00 ,40,40,40
BEGIN DESCRIPTION:
46
END DESCRIPTION:
#Sta/Elev= 12
   -12.2   47.63    -2.2   47.63    -1.8   48.13       0   48.13      .3   47.53
      .5   47.53     1.2   46.13     2.8   46.13     3.2   47.63     5.5   47.63
     6.3   46.83    16.3   46.83
#Mann= 3 , 0 , 0
   -12.2    .033       0       0    .033       0     3.2    .033       0
#XS Ineff= 2 , 0
               0   48.13     3.2           47.63
Permanent Ineff=
       F       F
Bank Sta=0,3.2
XS Rating Curve= 0
Exp/Cntr=.3,.1

Type RM Length L Ch R = 1 ,2260.00 ,10,10,10
BEGIN DESCRIPTION:
45.01
END DESCRIPTION:
#Sta/Elev= 12
   -13.7      46    -3.7      46    -2.2    46.8       0    46.8      .5    46.5
     1.2      45     2.4      45     3.2    46.2     3.7      47     5.5      47
     6.7    46.4    16.7    46.4
#Mann= 3 , 0 , 0
   -13.7    .033       0       0    .033       0     3.7    .033       0
#XS Ineff= 2 , 0
               0    46.8     3.7              47
Permanent Ineff=
       F       F
Bank Sta=0,3.7
XS Rating Curve= 0
Exp/Cntr=.3,.1

Type RM Length L Ch R = 1 ,2250.00 ,50,50,50
BEGIN DESCRIPTION:
45
END DESCRIPTION:
#Sta/Elev= 12
   -12.7   44.96    -2.7   44.96     -.8   46.46       0   46.46      .5   46.16
     1.2   44.66     2.4   44.66     3.2   45.86     3.7   46.66     5.5   46.66
     6.7   46.06    16.7   46.06
#Mann= 3 , 0 , 0
   -12.7    .033       0       0    .033       0     3.7    .033       0
#XS Ineff= 2 , 0
               0   46.46     3.7           46.66
Permanent Ineff=
       F       F
Bank Sta=0,3.7
XS Rating Curve= 0
Exp/Cntr=.3,.1

Type RM Length L Ch R = 1 ,2200.00 ,50,50,50
BEGIN DESCRIPTION:
44
END DESCRIPTION:
#Sta/Elev= 14
   -12.4   43.34    -2.4   43.34     -.8   44.84       0   44.84      .4   44.44
     1.1   43.04     1.9   43.04     2.3   43.44     2.9   43.64     3.4   44.54
     4.2   44.94       6   44.94     6.8   44.24    16.8   44.24
#Mann= 3 , 0 , 0
   -12.4    .033       0       0    .033       0     4.2    .033       0
#XS Ineff= 2 , 0
               0   44.84     4.2           44.94
Permanent Ineff=
       F       F
Bank Sta=0,4.2
XS Rating Curve= 0
Exp/Cntr=.3,.1

Type RM Length L Ch R = 1 ,2150.00 ,38,38,38
BEGIN DESCRIPTION:
43
END DESCRIPTION:
#Sta/Elev= 14
   -12.4   41.59    -2.4   41.59     -.8   43.09       0   43.09      .4   42.69
     1.1   41.99     1.9   41.99     2.3   42.39     2.9   42.59     3.5   43.49
     4.3   43.89     6.1   43.89     6.9   43.19    16.9   43.19
#Mann= 3 , 0 , 0
   -12.4    .033       0       0    .033       0     4.3    .033       0
#XS Ineff= 2 , 0
               0   43.09     4.3           43.89
Permanent Ineff=
       F       F
Bank Sta=0,4.3
XS Rating Curve= 0
Exp/Cntr=.3,.1

Type RM Length L Ch R = 1 ,2112.00 ,12,12,12
BEGIN DESCRIPTION:
42.012
END DESCRIPTION:
#Sta/Elev= 12
   -12.7   41.18    -2.7   41.18     -.8   42.68       0   42.68      .6   42.08
     1.6   41.28     2.6   41.08     3.4   42.28     4.1   42.98     5.6   42.98
     5.9   42.78    15.9   42.78
#Mann= 3 , 0 , 0
   -12.7    .033       0       0    .033       0     4.1    .033       0
#XS Ineff= 2 , 0
               0   42.68     4.1           42.98
Permanent Ineff=
       F       F
Bank Sta=0,4.1
XS Rating Curve= 0
Exp/Cntr=.3,.1

Type RM Length L Ch R = 1 ,2100.00 ,50,50,50
BEGIN DESCRIPTION:
42
END DESCRIPTION:
#Sta/Elev= 12
   -12.4   41.02    -2.4   41.02     -.8   42.52       0   42.52      .8   41.92
     1.6   40.92     3.4   40.92       4   42.02     4.8   42.62       7   42.62
      11   41.32      21   41.32
#Mann= 3 , 0 , 0
   -12.4    .033       0       0    .033       0     4.8    .033       0
#XS Ineff= 2 , 0
               0   42.52     4.8           42.62
Permanent Ineff=
       F       F
Bank Sta=0,4.8
XS Rating Curve= 0
Exp/Cntr=.3,.1

Type RM Length L Ch R = 1 ,2050.00 ,50,50,50
BEGIN DESCRIPTION:
41
END DESCRIPTION:
#Sta/Elev= 12
   -12.4   39.79    -2.4   39.79     -.8   41.29       0   41.29      .8   40.79
     1.6   39.69     3.4   39.69       4   40.89     4.8   41.49       7   41.49
      11   40.19      21   40.19
#Mann= 3 , 0 , 0
   -12.4    .033       0       0    .033       0     4.8    .033       0
#XS Ineff= 2 , 0
               0   41.29     4.8           41.49
Permanent Ineff=
       F       F
Bank Sta=0,4.8
XS Rating Curve= 0
Exp/Cntr=.3,.1

Type RM Length L Ch R = 1 ,2000.00 ,50,50,50
BEGIN DESCRIPTION:
40
END DESCRIPTION:
#Sta/Elev= 14
   -11.7   38.72    -1.7   38.72     -.5   40.12       0   40.12      .8   39.52
     1.6   38.52     2.6   38.52     2.8   38.92     3.6   38.92     3.9   39.52
     4.1   39.82     6.1   39.82     7.4   38.52    17.4   38.52
#Mann= 3 , 0 , 0
   -11.7    .033       0       0    .033       0     4.1    .033       0
#XS Ineff= 2 , 0
               0   40.12     4.1           39.82
Permanent Ineff=
       F       F
Bank Sta=0,4.1
XS Rating Curve= 0
Exp/Cntr=.3,.1

Type RM Length L Ch R = 1 ,1950.00 ,2,2,2
BEGIN DESCRIPTION:
39
END DESCRIPTION:
#Sta/Elev= 12
   -12.2   37.97    -2.2   37.97     -.6   38.57       0   38.77     1.4   37.07
     2.4   37.07     2.9   37.47     3.7   38.77     4.3   39.17     5.9   39.17
     7.9   37.57    17.9   37.57
#Mann= 3 , 0 , 0
   -12.2    .033       0       0    .033       0     4.3    .033       0
#XS Ineff= 2 , 0
               0   38.77     4.3           39.17
Permanent Ineff=
       F       F
Bank Sta=0,4.3
XS Rating Curve= 0
Exp/Cntr=.3,.1

Type RM Length L Ch R = 1 ,1948.00 ,48,48,48
BEGIN DESCRIPTION:
38.048
END DESCRIPTION:
#Sta/Elev= 12
   -12.2   37.84    -2.2   37.84     -.6   38.44       0   38.64     1.4   37.04
     2.4   37.04     2.9   37.44     3.7   38.74     4.3   39.14     5.9   39.14
     7.9   37.54    17.9   37.54
#Mann= 3 , 0 , 0
   -12.2    .033       0       0    .033       0     4.3    .033       0
#XS Ineff= 2 , 0
               0   38.64     4.3           39.14
Permanent Ineff=
       F       F
Bank Sta=0,4.3
XS Rating Curve= 0
Exp/Cntr=.3,.1

Type RM Length L Ch R = 1 ,1900.00 ,50,50,50
BEGIN DESCRIPTION:
38
END DESCRIPTION:
#Sta/Elev= 13
   -11.3   36.98    -1.3   36.98     -.6   37.68       0   37.68      .6   37.08
     1.1   36.78     2.1   36.38     3.1   36.18     3.7   37.28     4.5   37.78
     5.3   37.78     7.1   36.28    17.1   36.28
#Mann= 3 , 0 , 0
   -11.3    .033       0       0    .033       0     4.5    .033       0
#XS Ineff= 2 , 0
               0   37.68     4.5           37.78
Permanent Ineff=
       F       F
Bank Sta=0,4.5
XS Rating Curve= 0
Exp/Cntr=.3,.1

Type RM Length L Ch R = 1 ,1850.00 ,32,32,32
BEGIN DESCRIPTION:
37
END DESCRIPTION:
#Sta/Elev= 13
   -11.3   35.87    -1.3   35.87     -.6   36.57       0   36.57      .6   35.97
     1.1   35.57     2.1   35.07     3.1   34.97     3.7   36.07     4.5   36.57
     5.3   36.57     7.1   35.07    17.1   35.07
#Mann= 3 , 0 , 0
   -11.3    .033       0       0    .033       0     4.5    .033       0
#XS Ineff= 2 , 0
               0   36.57     4.5           36.57
Permanent Ineff=
       F       F
Bank Sta=0,4.5
XS Rating Curve= 0
Exp/Cntr=.3,.1

Type RM Length L Ch R = 1 ,1818.00 ,18,18,18
BEGIN DESCRIPTION:
36.018
END DESCRIPTION:
#Sta/Elev= 12
   -12.4   34.42    -2.4   34.42      -1   35.72       0   35.72      .4   35.32
     1.4   34.02       3   34.02     3.9   35.42     4.3   35.92     5.5   35.92
     6.1   35.32    16.1   35.32
#Mann= 3 , 0 , 0
   -12.4    .033       0       0    .033       0     4.3    .033       0
#XS Ineff= 2 , 0
               0   35.72     4.3           35.92
Permanent Ineff=
       F       F
Bank Sta=0,4.3
XS Rating Curve= 0
Exp/Cntr=.3,.1

Type RM Length L Ch R = 1 ,1800.00 ,50,50,50
BEGIN DESCRIPTION:
36
END DESCRIPTION:
#Sta/Elev= 12
   -12.4   34.18    -2.4   34.18      -1   35.48       0   35.48      .4   35.18
     1.4   33.88       3   33.88     3.9   35.28     4.3   35.78     5.5   35.78
     6.1   35.18    16.1   35.18
#Mann= 3 , 0 , 0
   -12.4    .033       0       0    .033       0     4.3    .033       0
#XS Ineff= 2 , 0
               0   35.48     4.3           35.78
Permanent Ineff=
       F       F
Bank Sta=0,4.3
XS Rating Curve= 0
Exp/Cntr=.3,.1

Type RM Length L Ch R = 1 ,1750.00 ,50,50,50
BEGIN DESCRIPTION:
35
END DESCRIPTION:
#Sta/Elev= 12
   -12.4   33.09    -2.4   33.09      -1   34.39       0   34.39      .4   33.99
     1.4   32.69       3   32.69     3.9   34.19     4.3   34.69     5.5   34.69
     6.1   34.09    16.1   34.09
#Mann= 3 , 0 , 0
   -12.4    .033       0       0    .033       0     4.3    .033       0
#XS Ineff= 2 , 0
               0   34.39     4.3           34.69
Permanent Ineff=
       F       F
Bank Sta=0,4.3
XS Rating Curve= 0
Exp/Cntr=.3,.1

Type RM Length L Ch R = 1 ,1700.00 ,50,50,50
BEGIN DESCRIPTION:
34
END DESCRIPTION:
#Sta/Elev= 14
   -11.8    31.9    -1.8    31.9     -.8      33       0      33      .8    32.4
     1.7    31.3     2.4    31.3     2.7    31.5     3.8    31.8     4.1    32.7
     5.9    33.7     6.3    33.7     6.6    33.4    16.6    33.4
#Mann= 3 , 0 , 0
   -11.8    .033       0       0    .033       0     5.9    .033       0
#XS Ineff= 2 , 0
               0      33     5.9            33.7
Permanent Ineff=
       F       F
Bank Sta=0,5.9
XS Rating Curve= 0
Exp/Cntr=.3,.1

Type RM Length L Ch R = 1 ,1650.00 ,13,13,13
BEGIN DESCRIPTION:
33
END DESCRIPTION:
#Sta/Elev= 11
   -15.3   31.21    -5.3   31.21    -4.7   32.31       0   32.31      .6   30.91
     3.1   30.91       4   32.21     6.2   33.81       7   33.81     7.3   33.51
    17.3   33.51
#Mann= 3 , 0 , 0
   -15.3    .033       0       0    .033       0     6.2    .033       0
#XS Ineff= 2 , 0
               0   32.31     6.2           33.81
Permanent Ineff=
       F       F
Bank Sta=0,6.2
XS Rating Curve= 0
Exp/Cntr=.3,.1

Type RM Length L Ch R = 1 ,1637.00 ,37,37,37
BEGIN DESCRIPTION:
32.037
END DESCRIPTION:
#Sta/Elev= 11
   -15.3    30.7    -5.3    30.7    -4.7    31.8       0    31.8      .6    30.8
     3.1    30.8       4    31.7     6.2    33.3       7    33.3     7.3    33.3
    17.3      33
#Mann= 3 , 0 , 0
   -15.3    .033       0       0    .033       0     6.2    .033       0
#XS Ineff= 2 , 0
               0    31.8     6.2            33.3
Permanent Ineff=
       F       F
Bank Sta=0,6.2
XS Rating Curve= 0
Exp/Cntr=.3,.1

Type RM Length L Ch R = 1 ,1600.00 ,42,42,42
BEGIN DESCRIPTION:
32
END DESCRIPTION:
#Sta/Elev= 12
   -14.9   30.56    -4.9   30.56    -4.1   31.26    -3.1   31.46       0   31.46
      .5   30.46      .8   30.46     1.4   30.16     2.4   30.16     3.2   31.46
     4.7   32.76    14.7   32.76
#Mann= 3 , 0 , 0
   -14.9    .033       0       0    .033       0     4.7    .033       0
#XS Ineff= 2 , 0
               0   31.46     4.7           32.76
Permanent Ineff=
       F       F
Bank Sta=0,4.7
XS Rating Curve= 0
Exp/Cntr=.3,.1

Type RM Length L Ch R = 1 ,1558.00 ,8,8,8
BEGIN DESCRIPTION:
31.008
END DESCRIPTION:
#Sta/Elev= 9
   -15.8   30.08    -5.8   30.08      -4   31.08       0   31.08      .4   29.48
     2.9   29.48     3.1   31.08     8.1   31.68    13.1   32.28
#Mann= 3 , 0 , 0
   -15.8    .033       0       0    .033       0     3.1    .033       0
#XS Ineff= 2 , 0
               0   31.08     3.1           31.08
Permanent Ineff=
       F       F
Bank Sta=0,3.1
XS Rating Curve= 0
Exp/Cntr=.3,.1

Type RM Length L Ch R = 1 ,1550.00 ,50,50,50
BEGIN DESCRIPTION:
31
END DESCRIPTION:
#Sta/Elev= 12
     -10    30.7       0    30.7      .7      30     1.2    29.3     1.8    29.3
       2      29     3.5      29     3.9    30.6     5.4    31.8     6.4    31.8
       8    32.5      18    32.5
#Mann= 3 , 0 , 0
     -10    .033       0       0    .033       0     5.4    .033       0
#XS Ineff= 2 , 0
               0    30.7     5.4            31.8
Permanent Ineff=
       F       F
Bank Sta=0,5.4
XS Rating Curve= 0
Exp/Cntr=.3,.1

Type RM Length L Ch R = 1 ,1500.00 ,50,50,50
BEGIN DESCRIPTION:
30
END DESCRIPTION:
#Sta/Elev= 14
     -13   28.57      -3   28.57      -1   29.77       0   29.77      .7   29.07
     1.2   28.37     1.8   28.37       2   27.97     3.5   27.97     3.9   29.67
     5.4   30.87     6.4   30.87       8   31.57      18   31.57
#Mann= 3 , 0 , 0
     -13    .033       0       0    .033       0     5.4    .033       0
#XS Ineff= 2 , 0
               0   29.77     5.4           30.87
Permanent Ineff=
       F       F
Bank Sta=0,5.4
XS Rating Curve= 0
Exp/Cntr=.3,.1

Type RM Length L Ch R = 1 ,1450.00 ,50,50,50
BEGIN DESCRIPTION:
29
END DESCRIPTION:
#Sta/Elev= 11
   -14.3   26.69    -4.3   26.69    -2.3   28.29       0   28.29      .6   27.89
     1.6   26.49     3.4   26.49     3.9   28.19     6.9   29.79     8.5   30.39
    18.5   30.39
#Mann= 3 , 0 , 0
   -14.3    .033       0       0    .033       0     8.5    .033       0
#XS Ineff= 2 , 0
               0   28.29     8.5           30.39
Permanent Ineff=
       F       F
Bank Sta=0,8.5
XS Rating Curve= 0
Exp/Cntr=.3,.1

Type RM Length L Ch R = 1 ,1400.00 ,7,7,7
BEGIN DESCRIPTION:
28
END DESCRIPTION:
#Sta/Elev= 11
   -14.3   25.22    -4.3   25.22    -2.3   26.82       0   26.82      .6   26.42
     1.6   25.02     3.4   25.02     3.9   26.72     6.9   28.32     8.5   28.92
    18.5   28.92
#Mann= 3 , 0 , 0
   -14.3    .033       0       0    .033       0     8.5    .033       0
#XS Ineff= 2 , 0
               0   26.82     8.5           28.92
Permanent Ineff=
       F       F
Bank Sta=0,8.5
XS Rating Curve= 0
Exp/Cntr=.3,.1

Type RM Length L Ch R = 1 ,1393.00 ,43,43,43
BEGIN DESCRIPTION:
27.043
END DESCRIPTION:
#Sta/Elev= 10
   -13.3   25.15    -3.3   25.15    -1.7   26.75       0   26.75      .4   26.15
     1.4   24.55     2.8   24.55     3.6   26.35     4.1   27.15    14.1   27.15
#Mann= 3 , 0 , 0
   -13.3    .033       0       0    .033       0     4.1    .033       0
#XS Ineff= 2 , 0
               0   26.75     4.1           27.15
Permanent Ineff=
       F       F
Bank Sta=0,4.1
XS Rating Curve= 0
Exp/Cntr=.3,.1

Type RM Length L Ch R = 1 ,1350.00 ,50,50,50
BEGIN DESCRIPTION:
27
END DESCRIPTION:
#Sta/Elev= 13
   -12.4   23.95    -2.4   23.95    -1.4   25.35     -.8   25.35     -.2   25.05
       0   25.05      .8   24.05     2.9   24.05     3.7   24.75     4.5   25.35
     5.3   25.35     6.3   24.75    16.3   24.75
#Mann= 3 , 0 , 0
   -12.4    .033       0     -.8    .033       0     4.5    .033       0
#XS Ineff= 2 , 0
             -.8   25.35     4.5           25.35
Permanent Ineff=
       F       F
Bank Sta=-.8,4.5
XS Rating Curve= 0
Exp/Cntr=.3,.1

Type RM Length L Ch R = 1 ,1300.00 ,50,50,50
BEGIN DESCRIPTION:
26
END DESCRIPTION:
#Sta/Elev= 15
   -12.4   23.37    -2.4   23.37    -1.4   24.77     -.8   24.77     -.2   24.47
       0   24.47      .8   23.47     2.2   23.47     2.4   23.17     3.1   23.17
     3.9   23.87     4.7   24.47     5.5   24.47     6.5   23.87    16.5   23.87
#Mann= 3 , 0 , 0
   -12.4    .033       0       0    .033       0     4.7    .033       0
#XS Ineff= 2 , 0
               0   24.47     4.7           24.47
Permanent Ineff=
       F       F
Bank Sta=0,4.7
XS Rating Curve= 0
Exp/Cntr=.3,.1

Type RM Length L Ch R = 1 ,1250.00 ,50,50,50
BEGIN DESCRIPTION:
25
END DESCRIPTION:
#Sta/Elev= 15
   -12.4   22.36    -2.4   22.36    -1.4   23.76     -.8   23.76     -.2   23.46
       0   23.46      .8   22.06     2.2   22.06     2.4   22.76     3.1   22.76
     3.9   23.46     4.7   24.06     5.5   24.06     6.5   23.46    16.5   23.46
#Mann= 3 , 0 , 0
   -12.4    .033       0       0    .033       0     4.7    .033       0
#XS Ineff= 2 , 0
               0   23.46     4.7           24.06
Permanent Ineff=
       F       F
Bank Sta=0,4.7
XS Rating Curve= 0
Exp/Cntr=.3,.1

Type RM Length L Ch R = 1 ,1200.00 ,50,50,50
BEGIN DESCRIPTION:
24
END DESCRIPTION:
#Sta/Elev= 15
   -13.7    21.6    -3.7    21.6    -1.9    23.1    -1.2    23.1     -.4    22.7
       0    22.7      .6    21.3      .6      21     2.1      21     2.1    21.3
     2.3    21.3     2.9    22.8     3.5    22.8     5.1    23.6    15.1    23.6
#Mann= 3 , 0 , 0
   -13.7    .033       0       0    .033       0     2.9    .033       0
#XS Ineff= 2 , 0
               0    22.7     2.9            22.8
Permanent Ineff=
       F       F
Bank Sta=0,2.9
XS Rating Curve= 0
Exp/Cntr=.3,.1

Type RM Length L Ch R = 1 ,1150.00 ,50,50,50
BEGIN DESCRIPTION:
23
END DESCRIPTION:
#Sta/Elev= 19
   -13.7   20.63    -3.7   20.63    -2.2   21.93    -1.3   21.93     -.3   21.63
       0   21.63      .5   20.33     .65   20.33     .65   20.18    1.35   20.18
    1.95   20.58    2.45   20.58    2.85   21.48    3.45   21.48    6.45   22.88
    7.85   23.48    8.25   23.48    8.55   23.28   18.55   23.28
#Mann= 3 , 0 , 0
   -13.7    .033       0       0    .033       0    7.85    .033       0
#XS Ineff= 2 , 0
               0   21.63    7.85           23.48
Permanent Ineff=
       F       F
Bank Sta=0,7.85
XS Rating Curve= 0
Exp/Cntr=.3,.1

Type RM Length L Ch R = 1 ,1100.00 ,50,50,50
BEGIN DESCRIPTION:
22
END DESCRIPTION:
#Sta/Elev= 19
   -13.7   19.88    -3.7   19.88    -2.2   21.18    -1.3   21.18     -.3   20.88
       0   20.88      .5   19.58     .65   19.58     .65   19.43    1.35   19.43
    1.95   19.83    2.45   19.83    2.85   20.73    3.45   20.73    6.45   22.13
    7.85   22.73    8.25   22.73    8.55   22.53   18.55   22.53
#Mann= 3 , 0 , 0
   -13.7    .033       0       0    .033       0    7.85    .033       0
#XS Ineff= 2 , 0
               0   20.88    7.85           22.73
Permanent Ineff=
       F       F
Bank Sta=0,7.85
XS Rating Curve= 0
Exp/Cntr=.3,.1

Type RM Length L Ch R = 1 ,1050.00 ,50,50,50
BEGIN DESCRIPTION:
21
END DESCRIPTION:
#Sta/Elev= 11
   -13.6   19.39    -3.6   19.39    -2.2   20.59    -1.4   20.59     -.8   20.19
       0   20.19      .3   19.19     1.3   18.79     3.3   18.79     3.8   20.39
    13.8   20.39
#Mann= 3 , 0 , 0
   -13.6    .033       0       0    .033       0     3.8    .033       0
#XS Ineff= 2 , 0
               0   20.19     3.8           20.39
Permanent Ineff=
       F       F
Bank Sta=0,3.8
XS Rating Curve= 0
Exp/Cntr=.3,.1

Type RM Length L Ch R = 1 ,1000.00 ,6,6,6
BEGIN DESCRIPTION:
20
END DESCRIPTION:
#Sta/Elev= 11
   -13.6    18.7    -3.6    18.7    -2.2    19.9    -1.4    19.9     -.8    19.5
       0    19.5      .3      19     1.3    18.7     3.3    18.4     3.8    19.4
    13.8    19.4
#Mann= 3 , 0 , 0
   -13.6    .033       0       0    .033       0     3.8    .033       0
#XS Ineff= 2 , 0
               0    19.5     3.8            19.4
Permanent Ineff=
       F       F
Bank Sta=0,3.8
XS Rating Curve= 0
Exp/Cntr=.3,.1

Type RM Length L Ch R = 1 ,994.00  ,20,20,20
BEGIN DESCRIPTION:
19.044
END DESCRIPTION:
#Sta/Elev= 8
   -13.4   19.82    -3.4   19.82      -1   19.82       0   19.52      .4   18.02
     2.4   18.02     2.8   19.32    12.8   19.32
#Mann= 3 , 0 , 0
   -13.4    .015       0       0    .015       0     2.8    .015       0
#XS Ineff= 2 , 0
               0   19.52     2.8           19.32
Permanent Ineff=
       F       F
Bank Sta=0,2.8
XS Rating Curve= 0
Exp/Cntr=.3,.1

Type RM Length L Ch R = 1 ,974.00  ,24,24,24
BEGIN DESCRIPTION:
19.024
END DESCRIPTION:
#Sta/Elev= 16
   -10.6   19.76     -.6   19.76       0   19.46      .2   17.86       3   17.86
       3   19.36     3.2   19.36     3.2   17.86     4.8   17.86     4.8   19.36
       5   19.36       5   17.86      10   17.86      10   18.86    10.5   19.36
    20.5   19.36
#Mann= 3 , 0 , 0
   -10.6    .015       0       0    .015       0    10.5    .015       0
#XS Ineff= 2 , 0
               0   19.46    10.5           19.36
Permanent Ineff=
       F       F
Bank Sta=0,10.5
XS Rating Curve= 0
Exp/Cntr=.3,.1

Type RM Length L Ch R = 1 ,950.00  ,50,50,50
BEGIN DESCRIPTION:
19
END DESCRIPTION:
#Sta/Elev= 15
     -13   18.26      -3   18.26    -2.4   18.86     -.2   18.86     -.2   19.16
       0   19.16       0   18.06      .2   17.76     1.9   17.76     2.1   18.06
     2.1   19.06     2.3   19.06     4.8   19.06     6.1   17.66    16.1   17.66
#Mann= 3 , 0 , 0
     -13    .015       0       0    .015       0     2.1    .015       0
#XS Ineff= 2 , 0
               0   19.16     2.1           19.06
Permanent Ineff=
       F       F
Bank Sta=0,2.1
XS Rating Curve= 0
Exp/Cntr=.3,.1

Type RM Length L Ch R = 1 ,900.00  ,50,50,50
BEGIN DESCRIPTION:
18
END DESCRIPTION:
#Sta/Elev= 15
     -13   17.64      -3   17.64    -2.4   18.24     -.2   18.24     -.2   18.54
       0   18.54       0   17.74      .2   17.54     1.9   17.54     2.1   17.74
     2.1   18.74     2.3   18.74     4.8   18.74     6.1   17.34    16.1   17.34
#Mann= 3 , 0 , 0
     -13    .015       0       0    .015       0     2.1    .015       0
#XS Ineff= 2 , 0
               0   18.54     2.1           18.74
Permanent Ineff=
       F       F
Bank Sta=0,2.1
XS Rating Curve= 0
Exp/Cntr=.3,.1

Type RM Length L Ch R = 1 ,850.00  ,24,24,24
BEGIN DESCRIPTION:
17
END DESCRIPTION:
#Sta/Elev= 15
     -13    17.8      -3    17.8    -2.4    18.4     -.2    18.4     -.2    18.7
       0    18.7       0    17.3      .2    17.1     1.9    17.1     2.1    17.3
     2.1    18.9     2.3    18.9     4.8    18.9     6.1    17.5    16.1    17.5
#Mann= 3 , 0 , 0
     -13    .015       0       0    .015       0     2.1    .015       0
#XS Ineff= 2 , 0
               0    18.7     2.1            18.9
Permanent Ineff=
       F       F
Bank Sta=0,2.1
XS Rating Curve= 0
Exp/Cntr=.3,.1

Type RM Length L Ch R = 1 ,826.00  ,179,179,179
BEGIN DESCRIPTION:
16.026
END DESCRIPTION:
#Sta/Elev= 10
   -12.2   18.18    -2.2   18.18    -1.5   18.78       0   18.78      .6   18.18
      .6   16.18     2.6   16.18     2.6   18.18       3   18.58      13   18.58
#Mann= 3 , 0 , 0
   -12.2    .015       0       0    .015       0       3    .015       0
#XS Ineff= 2 , 0
               0   18.78       3           18.58
Permanent Ineff=
       F       F
Bank Sta=0,3
XS Rating Curve= 0
Exp/Cntr=.3,.1

Type RM Length L Ch R = 1 ,647.00  ,47,47,47
BEGIN DESCRIPTION:
12.047
END DESCRIPTION:
#Sta/Elev= 12
     -14   14.67      -4   14.67    -3.4   15.07       0   15.07      .2   15.07
      .2   13.77      .5   13.47     2.4   13.47     2.7   13.77     2.7   15.07
     4.9   15.87    14.9   15.87
#Mann= 3 , 0 , 0
     -14    .015       0       0    .015       0     4.9    .015       0
#XS Ineff= 2 , 0
               0   15.07     4.9           15.87
Permanent Ineff=
       F       F
Bank Sta=0,4.9
XS Rating Curve= 0
Exp/Cntr=.3,.1

Type RM Length L Ch R = 1 ,600.00  ,50,50,50
BEGIN DESCRIPTION:
12
END DESCRIPTION:
#Sta/Elev= 14
   -12.2   14.58    -2.2   14.58    -1.5   15.08       0   15.08     1.3   14.58
     1.5   14.58     1.5   13.38     1.8   13.08     3.7   13.08       4   13.38
       4   14.68       5   14.68     6.4   15.88    16.4   15.88
#Mann= 3 , 0 , 0
   -12.2    .015       0       0    .015       0       4    .015       0
#XS Ineff= 2 , 0
               0   15.08       4           14.68
Permanent Ineff=
       F       F
Bank Sta=0,4
XS Rating Curve= 0
Exp/Cntr=.3,.1

Type RM Length L Ch R = 1 ,550.00  ,26,26,26
BEGIN DESCRIPTION:
11
END DESCRIPTION:
#Sta/Elev= 13
   -12.2   13.92    -2.2   13.92    -1.5   14.42       0   14.42     1.3   13.82
     1.5   13.82     1.5   12.52     3.7   12.52       4   12.82       4   14.12
       5   14.12     6.4   15.32    16.4   15.32
#Mann= 3 , 0 , 0
   -12.2    .015       0       0    .015       0       4    .015       0
#XS Ineff= 2 , 0
               0   14.42       4           14.12
Permanent Ineff=
       F       F
Bank Sta=0,4
XS Rating Curve= 0
Exp/Cntr=.3,.1

Type RM Length L Ch R = 1 ,524.00  ,9,9,9
BEGIN DESCRIPTION:
10.024
END DESCRIPTION:
#Sta/Elev= 11
     -10   14.08       0   14.08       0   12.68      .3   12.28     2.2   12.28
     2.5   12.68     2.5   13.98     3.3   13.98     3.3   16.13     5.1   16.13
     5.1   18.13
#Mann= 3 , 0 , 0
     -10    .015       0       0    .015       0     2.5    .015       0
#XS Ineff= 2 , 0
               0   14.08     2.5           13.98
Permanent Ineff=
       F       F
Bank Sta=0,2.5
XS Rating Curve= 0
Exp/Cntr=.3,.1

Type RM Length L Ch R = 1 ,515.00  ,15,15,15
BEGIN DESCRIPTION:
10.015
END DESCRIPTION:
#Sta/Elev= 11
     -10    14.3       0    14.3       0    12.5      .3    12.1     2.2    12.1
     2.5    12.5     2.5    14.2     3.3    14.2     3.3   16.35     5.1   16.35
     5.1   18.35
#Mann= 3 , 0 , 0
     -10    .015       0       0    .015       0     2.5    .015       0
#XS Ineff= 2 , 0
               0    14.3     2.5            14.2
Permanent Ineff=
       F       F
Bank Sta=0,2.5
XS Rating Curve= 0
Exp/Cntr=.3,.1

Type RM Length L Ch R = 1 ,500.00  ,8,8,8
BEGIN DESCRIPTION:
10
END DESCRIPTION:
#Sta/Elev= 11
     -10   13.68       0   13.68       0   12.38      .3   12.08     2.2   12.08
     2.5   12.38     2.5   13.68     3.3   13.68     3.3   15.38     5.1   15.83
     5.1   17.83
#Mann= 3 , 0 , 0
     -10    .015       0       0    .015       0     2.5    .015       0
#XS Ineff= 2 , 0
               0   13.68     2.5           13.68
Permanent Ineff=
       F       F
Bank Sta=0,2.5
XS Rating Curve= 0
Exp/Cntr=.3,.1

Type RM Length L Ch R = 1 ,492.00  ,1,1,1
BEGIN DESCRIPTION:
9.042
END DESCRIPTION:
#Sta/Elev= 12
   -12.9   13.77    -2.9   13.77    -1.4   11.87     -.2   11.87     -.2   13.37
       0   13.37       0   11.97     2.5   11.97     2.5   13.37     3.3   13.37
     3.3   15.37    13.3   15.37
#Mann= 3 , 0 , 0
   -12.9    .015       0       0    .015       0     2.5    .015       0
#XS Ineff= 2 , 0
               0   13.37     2.5           13.37
Permanent Ineff=
       F       F
Bank Sta=0,2.5
XS Rating Curve= 0
Exp/Cntr=.3,.1

Type RM Length L Ch R = 1 ,491.00  ,9,9,9
BEGIN DESCRIPTION:
9.041
END DESCRIPTION:
#Sta/Elev= 14
   -12.9   13.77    -2.9   13.77    -1.4   11.87     -.2   11.87     -.2   13.37
       0   13.37       0   11.97       0   11.07     2.5   11.07     2.5   11.97
     2.5   13.37     3.3   13.37     3.3   15.37    13.3   15.37
#Mann= 3 , 0 , 0
   -12.9    .015       0       0    .015       0     2.5    .015       0
#XS Ineff= 2 , 0
               0   13.37     2.5           13.37
Permanent Ineff=
       F       F
Bank Sta=0,2.5
XS Rating Curve= 0
Exp/Cntr=.3,.1

Type RM Length L Ch R = 1 ,482.00  ,32,32,32
BEGIN DESCRIPTION:
9.032
END DESCRIPTION:
#Sta/Elev= 18
     -10   13.23       0   13.23      .8   13.23      .8   12.68     1.3   12.68
     1.3   11.58     1.6    9.98     1.8    9.98     1.8    9.68     4.8    9.68
     4.8    9.98       5    9.98     5.3   11.58     5.3   12.68     5.8   12.68
     5.8   13.23     6.6   13.23    16.6   13.23
#Mann= 3 , 0 , 0
     -10    .015       0      .8    .015       0     5.8    .015       0
#XS Ineff= 2 , 0
              .8   13.23     5.8           13.23
Permanent Ineff=
       F       F
Bank Sta=.8,5.8
XS Rating Curve= 0
Exp/Cntr=.3,.1

Type RM Length L Ch R = 1 ,450.00  ,50,50,50
BEGIN DESCRIPTION:
9
END DESCRIPTION:
#Sta/Elev= 10
     -13   12.21      -3   12.21    -2.2   12.81       0   12.81      .5   11.31
       5   11.31     5.5   12.71     7.8   12.71     8.3   12.31    18.3   12.31
#Mann= 3 , 0 , 0
     -13    .015       0       0    .015       0     5.5    .015       0
#XS Ineff= 2 , 0
               0   12.81     5.5           12.71
Permanent Ineff=
       F       F
Bank Sta=0,5.5
XS Rating Curve= 0
Exp/Cntr=.3,.1

Type RM Length L Ch R = 1 ,400.00  ,6,6,6
BEGIN DESCRIPTION:
8
END DESCRIPTION:
#Sta/Elev= 10
     -13   12.25      -3   12.25    -2.2   12.85       0   12.85      .5   11.05
       5   11.05     5.5   12.75     7.8   12.75     8.3   12.35    18.3   12.35
#Mann= 3 , 0 , 0
     -13    .033       0       0    .033       0     5.5    .033       0
#XS Ineff= 2 , 0
               0   12.85     5.5           12.75
Permanent Ineff=
       F       F
Bank Sta=0,5.5
XS Rating Curve= 0
Exp/Cntr=.3,.1

Type RM Length L Ch R = 1 ,394.00  ,44,44,44
BEGIN DESCRIPTION:
7.044
END DESCRIPTION:
#Sta/Elev= 10
     -13   12.01      -3   12.01    -2.2   12.61       0   12.61      .5   11.01
       5   11.01     5.5   12.51     7.8   12.51     8.3   12.11    18.3   12.11
#Mann= 3 , 0 , 0
     -13    .033       0       0    .033       0     5.5    .033       0
#XS Ineff= 2 , 0
               0   12.61     5.5           12.51
Permanent Ineff=
       F       F
Bank Sta=0,5.5
XS Rating Curve= 0
Exp/Cntr=.3,.1

Type RM Length L Ch R = 1 ,350.00  ,50,50,50
BEGIN DESCRIPTION:
7
END DESCRIPTION:
#Sta/Elev= 10
     -13   11.72      -3   11.72    -2.2   12.31       0   12.32      .5   10.62
       5   10.62     5.5   12.22     7.8   12.22     8.3   11.82    18.3   11.82
#Mann= 3 , 0 , 0
     -13    .033       0       0    .033       0     5.5    .033       0
#XS Ineff= 2 , 0
               0   12.32     5.5           12.22
Permanent Ineff=
       F       F
Bank Sta=0,5.5
XS Rating Curve= 0
Exp/Cntr=.3,.1

Type RM Length L Ch R = 1 ,300.00  ,50,50,50
BEGIN DESCRIPTION:
6
END DESCRIPTION:
#Sta/Elev= 13
   -12.2   10.81    -2.2   10.81      -1   12.01       0   12.01       1   11.41
     1.2   10.61     6.7   10.61     7.1   10.11     7.8   10.11     8.2   11.21
    10.7   11.21    11.2   10.81    21.2   10.81
#Mann= 3 , 0 , 0
   -12.2    .033       0       0    .033       0     8.2    .033       0
#XS Ineff= 2 , 0
               0   12.01     8.2           11.21
Permanent Ineff=
       F       F
Bank Sta=0,8.2
XS Rating Curve= 0
Exp/Cntr=.3,.1

Type RM Length L Ch R = 1 ,250.00  ,50,50,50
BEGIN DESCRIPTION:
5
END DESCRIPTION:
#Sta/Elev= 14
   -14.3    10.3    -4.3    10.3    -3.1    11.5     -.6    11.7       0    11.7
      .3     9.7     1.2     9.5     5.3     9.5     5.8     9.9     6.2    11.6
     6.8    11.6     8.8    11.6     9.6    10.8    19.6    10.8
#Mann= 3 , 0 , 0
   -14.3    .033       0       0    .033       0     6.2    .033       0
#XS Ineff= 2 , 0
               0    11.7     6.2            11.6
Permanent Ineff=
       F       F
Bank Sta=0,6.2
XS Rating Curve= 0
Exp/Cntr=.3,.1

Type RM Length L Ch R = 1 ,200.00  ,50,50,50
BEGIN DESCRIPTION:
4
END DESCRIPTION:
#Sta/Elev= 14
   -14.3    9.94    -4.3    9.94    -3.1   11.14     -.6   11.34       0   11.34
      .3    9.34     1.2    9.14     5.3    9.14     5.8    9.54     6.2   11.24
     6.8   11.24     8.8   11.24     9.6   10.44    19.6   10.44
#Mann= 3 , 0 , 0
   -14.3    .033       0       0    .033       0     6.2    .033       0
#XS Ineff= 2 , 0
               0   11.34     6.2           11.24
Permanent Ineff=
       F       F
Bank Sta=0,6.2
XS Rating Curve= 0
Exp/Cntr=.3,.1

Type RM Length L Ch R = 1 ,150.00  ,36,36,36
BEGIN DESCRIPTION:
3
END DESCRIPTION:
#Sta/Elev= 13
   -14.3    9.78    -4.3    9.78    -3.1   10.98     -.6   11.18       0   11.18
     1.2    8.98     5.3    8.98     5.8    9.38     6.2   11.08     6.8   11.08
     8.8   11.08     9.6   10.28    19.6   10.28
#Mann= 3 , 0 , 0
   -14.3    .033       0       0    .033       0     6.2    .033       0
#XS Ineff= 2 , 0
               0   11.18     6.2           11.08
Permanent Ineff=
       F       F
Bank Sta=0,6.2
XS Rating Curve= 0
Exp/Cntr=.3,.1

Type RM Length L Ch R = 1 ,114.00  ,12,12,12
BEGIN DESCRIPTION:
2.014
END DESCRIPTION:
#Sta/Elev= 12
   -14.3    9.29    -4.3    9.29      -3   10.29     -.6   11.09       0   11.09
      .3    8.59     6.3    8.59     6.3   10.79     6.6   11.09     9.4   11.09
    10.7    9.99    20.7    9.99
#Mann= 3 , 0 , 0
   -14.3    .033       0       0    .033       0     6.6    .033       0
#XS Ineff= 2 , 0
               0   11.09     6.6           11.09
Permanent Ineff=
       F       F
Bank Sta=0,6.6
XS Rating Curve= 0
Exp/Cntr=.3,.1

Type RM Length L Ch R = 1 ,102.00  ,2,2,2
BEGIN DESCRIPTION:
2.002
END DESCRIPTION:
#Sta/Elev= 15
   -13.1    9.41    -3.1    9.41    -1.1   10.61     -.6   10.61       0   10.61
      .3    9.41     3.2    9.41     3.2    8.71    5.55    8.71    5.55    9.41
     8.3    9.41     8.5   10.61    10.8   10.61    12.3    9.21    22.3    9.21
#Mann= 3 , 0 , 0
   -13.1    .033       0       0    .033       0     8.5    .033       0
#XS Ineff= 2 , 0
               0   10.61     8.5           10.61
Permanent Ineff=
       F       F
Bank Sta=0,8.5
XS Rating Curve= 0
Exp/Cntr=.3,.1

Type RM Length L Ch R = 1 ,100.00  ,50,50,50
BEGIN DESCRIPTION:
2
END DESCRIPTION:
#Sta/Elev= 11
   -13.1    9.41    -3.1    9.41    -1.1   10.61     -.6   10.61       0   10.61
      .4    8.61     8.4    8.61     8.6   10.31    10.9   10.31    12.4    8.91
    22.4    8.91
#Mann= 3 , 0 , 0
   -13.1    .033       0       0    .033       0     8.6    .033       0
#XS Ineff= 2 , 0
               0   10.61     8.6           10.31
Permanent Ineff=
       F       F
Bank Sta=0,8.6
XS Rating Curve= 0
Exp/Cntr=.3,.1

Type RM Length L Ch R = 1 ,50.00   ,44,44,44
BEGIN DESCRIPTION:
1
END DESCRIPTION:
#Sta/Elev= 11
   -13.1    8.84    -3.1    8.84    -1.1   10.04     -.6   10.04       0   10.04
      .4    7.94     8.4    7.94     8.6    9.74    10.9    9.74    12.4    8.34
    22.4    8.34
#Mann= 3 , 0 , 0
   -13.1    .033       0       0    .033       0     8.6    .033       0
#XS Ineff= 2 , 0
               0   10.04     8.6            9.74
Permanent Ineff=
       F       F
Bank Sta=0,8.6
XS Rating Curve= 0
Exp/Cntr=.3,.1

Type RM Length L Ch R = 1 ,6.00    ,6,6,6
BEGIN DESCRIPTION:
0.006
END DESCRIPTION:
#Sta/Elev= 15
   -19.7   10.03    -9.7   10.03    -8.2   10.73    -2.7   10.73     -.6    9.63
       0    9.63       0    7.23    11.4    7.23    11.7    9.53    12.3    9.53
    14.5    9.53    16.7   11.33    20.7   11.33    24.2    8.93    34.2    8.93
#Mann= 3 , 0 , 0
   -19.7    .033       0       0    .033       0    11.7    .033       0
#XS Ineff= 2 , 0
               0    9.63    11.7            9.53
Permanent Ineff=
       F       F
Bank Sta=0,11.7
XS Rating Curve= 0
Exp/Cntr=.3,.1

Type RM Length L Ch R = 1 ,0.00    ,0,0,0
BEGIN DESCRIPTION:
0
END DESCRIPTION:
#Sta/Elev= 6
     -10   11.18       0   11.18       0    7.18    11.5    7.18    11.5   11.18
    21.5   11.18
#Mann= 3 , 0 , 0
     -10    .033       0       0    .033       0    11.5    .033       0
#XS Ineff= 2 , 0
               0   11.18    11.5           11.18
Permanent Ineff=
       F       F
Bank Sta=0,11.5
XS Rating Curve= 0
Exp/Cntr=.3,.1

Chan Stop Cuts=-1
