--- DONGSIL.prj (project) ---

Proj Title=DONGSIL
Current Plan=p01
Default Exp/Contr=.3,.1
SI Units
Geom File=g01
Flow File=f01
Plan File=p01
Y Axis Title=Elevation
X Axis Title(PF)=Main Channel Distance
X Axis Title(XS)=Station
BEGIN DESCRIPTION:
           BACK WATER COMPUTATION
      APPLICATION OF HEC-2 BY Samju Construction Engineering
      DONGSIL-STREEM : 30 YR
END DESCRIPTION:
DSS Export Rating Curves= 0
DSS Export Rating Curve Sorted= 0
DSS Export Volume Flow Curves= 0
DXF OffsetX= 0
DXF OffsetY= 0
DXF ScaleX= 1
DXF ScaleY= 10

--- DONGSIL.p01 (plan) ---

Plan Title=Imported Plan 01
Version=Version 3.0.1  Mar 2001
Short Identifier=Imported Pla
Geom File=g01
Flow File=f01
Subcritical Flow
K Sum by GR= 0
Std Step Tol= 0.003
Critical Tol= 0.003
Num of Std Step Trials= 20
Max Error Tol= 0.1
Flow Tol Ratio= 0.001
Split Flow NTrial= 30
Split Flow Tol= 0.02
Split Flow Ratio= 0.02
Log Output Level= 0
Friction Slope Method= 1
Unsteady Friction Slope Method= 2
Parabolic Critical Depth
Global Vel Dist= 0 , 0 , 0
Global Log Level= 0
CheckData=True
Encroach Param=-1 ,0,0, 0
Computation Interval=1HOUR
Output Interval=1HOUR
Run HTab= 0
Run UNet= 0
Run PostProcess= 0
UNET Theta= 1
UNET ZTol= 0.02
UNET ZSATol= 0.1
UNET MxIter= 20
UNET MaxInSteps= 20
UNET DtIC= 0
UNET DtMin= 0
UNET MaxCRTS= 20
UNET WFStab= 2
UNET SFStab= 1
UNET WFX= 1
UNET SFX= 1
UNET Convert EG Bridges=-1
UNET Use Existing IB Tables=-1
Instantaneous Interval=1HOUR
Write IC File= 0
Write Velocity= 0
Write Detailed= 0

--- DONGSIL.f01 (steady flow) ---

Flow Title=Imported Flow 01
Version=Version 3.0.1  Mar 2001
Number of Profiles= 1
Profile Names=PF 1
River Rch & RM=RIVER-1,Reach-1         ,72.015
      75
Boundary for River Rch & Prof#=RIVER-1,Reach-1         , 1
Up Type= 0
Dn Type= 3
Dn Slope=.0109
DSS Import GetInterval= 0
DSS Import GetPeak= 0
DSS Import FillOption= 0

--- DONGSIL.g01 (geometry) ---

Geom Title=Imported Geom 01
Version=Version 3.0.1  Mar 2001

River Reach=RIVER-1         ,Reach-1
Reach XY= 2
              .5             .95              .5             .05

Type RM Length L Ch R = 1 ,72.015  ,15,15,15
#Sta/Elev= 12
    -6.7   92.63    -4.7   91.13    -2.7   89.63     -.7   88.13       0   87.23
       1   86.03     1.7   86.03     2.5   86.33     3.4   87.23     4.2   87.23
     6.2   86.33    16.2   86.33
#Mann= 3 , 0 , 0
    -6.7    .033       0       0    .033       0     3.4    .033       0
Bank Sta=0,3.4
XS Rating Curve= 0
Exp/Cntr=.3,.1

Type RM Length L Ch R = 1 ,72      ,29,29,29
#Sta/Elev= 13
   -10.5   91.04    -5.5   89.04     -.5   87.04       0   86.04     1.2   85.34
     1.6   84.74     2.6   84.74     2.9   84.94     3.7   85.04     4.1   85.74
     4.4   85.74     5.1   85.24    15.1   85.24
#Mann= 3 , 0 , 0
   -10.5    .033       0       0    .033       0     4.1    .033       0
Bank Sta=0,4.1
XS Rating Curve= 0
Exp/Cntr=.3,.1

Type RM Length L Ch R = 1 ,71.021  ,21,21,21
#Sta/Elev= 7
     -10   85.99       0   85.99      .6   85.39     1.4   85.39     2.2   85.99
     7.2   86.79    12.2   87.59
#Mann= 3 , 0 , 0
     -10    .033       0       0    .033       0     2.2    .033       0
Bank Sta=0,2.2
XS Rating Curve= 0
Exp/Cntr=.3,.1

Type RM Length L Ch R = 1 ,71      ,50,50,50
#Sta/Elev= 8
   -13.3   82.28    -3.3   82.28    -3.3   83.78       0   83.78      .8   83.08
     1.7   83.08     2.9   84.58    12.9   84.58
#Mann= 3 , 0 , 0
   -13.3    .033       0       0    .033       0     2.9    .033       0
Bank Sta=0,2.9
XS Rating Curve= 0
Exp/Cntr=.3,.1

Type RM Length L Ch R = 1 ,70      ,50,50,50
#Sta/Elev= 8
   -13.3    78.2    -3.3    78.2    -3.3    79.7       0    79.7      .8      79
     1.7      79     2.9    80.5    12.9    80.5
#Mann= 3 , 0 , 0
   -13.3    .033       0       0    .033       0     2.9    .033       0
Bank Sta=0,2.9
XS Rating Curve= 0
Exp/Cntr=.3,.1

Type RM Length L Ch R = 1 ,69      ,3,3,3
#Sta/Elev= 7
     -10   76.35       0   76.35      .7   75.45     1.9   75.45     2.6   76.35
     5.2   76.35     5.2   78.35
#Mann= 3 , 0 , 0
     -10    .033       0       0    .033       0     2.6    .033       0
Bank Sta=0,2.6
XS Rating Curve= 0
Exp/Cntr=.3,.1

Type RM Length L Ch R = 1 ,68.047  ,34,34,34
#Sta/Elev= 7
     -10   76.04       0   76.04      .7   75.04     1.9   75.04     2.6   76.04
     5.2   76.04     5.2   78.04
#Mann= 3 , 0 , 0
     -10    .033       0       0    .033       0     2.6    .033       0
Bank Sta=0,2.6
XS Rating Curve= 0
Exp/Cntr=.3,.1

Type RM Length L Ch R = 1 ,68.013  ,13,13,13
#Sta/Elev= 8
   -14.5   73.08    -4.5   73.08      -2   74.78       0   74.78      .3   73.48
       2   73.48     2.3   74.98    12.3   74.98
#Mann= 3 , 0 , 0
   -14.5    .033       0       0    .033       0     2.3    .033       0
Bank Sta=0,2.3
XS Rating Curve= 0
Exp/Cntr=.3,.1

Type RM Length L Ch R = 1 ,68      ,50,50,50
#Sta/Elev= 9
   -12.4   74.45    -2.4   74.45    -1.6   73.45       0   73.45     1.1   72.65
     1.9   72.65     2.7   73.35     3.7   73.35     3.7   74.85
#Mann= 3 , 0 , 0
   -12.4    .033       0       0    .033       0     2.7    .033       0
Bank Sta=0,2.7
XS Rating Curve= 0
Exp/Cntr=.3,.1

Type RM Length L Ch R = 1 ,67      ,41,41,41
#Sta/Elev= 13
     -15   72.16      -5   72.16    -4.7   72.46      -4   72.46      -3   71.66
      -1   70.36       0   70.06     1.6   68.56     3.7   68.56     5.7   70.16
     6.5   70.16     7.8   68.96    17.8   68.96
#Mann= 3 , 0 , 0
     -15    .033       0      -4    .033       0     5.7    .033       0
Bank Sta=-4,5.7
XS Rating Curve= 0
Exp/Cntr=.3,.1

Type RM Length L Ch R = 1 ,66.009  ,9,9,9
#Sta/Elev= 13
     -15    69.5      -5    69.5    -4.7    69.8      -4    69.8      -3      69
      -1    67.7       0    67.4     1.6    65.8     3.7    65.8     5.7    67.5
     6.5    67.5     7.8    66.3    17.8    66.3
#Mann= 3 , 0 , 0
     -15    .033       0      -4    .033       0     5.7    .033       0
Bank Sta=-4,5.7
XS Rating Curve= 0
Exp/Cntr=.3,.1

Type RM Length L Ch R = 1 ,66      ,43,43,43
#Sta/Elev= 13
     -14   68.87      -4   68.87    -3.7   69.17      -3   69.17      -2   68.37
       0   67.07       1   66.77     2.6   65.77     4.7   65.77     6.7   66.87
     7.5   66.87     8.8   65.67    18.8   65.67
#Mann= 3 , 0 , 0
     -14    .033       0      -3    .033       0     6.7    .033       0
Bank Sta=-3,6.7
XS Rating Curve= 0
Exp/Cntr=.3,.1

Type RM Length L Ch R = 1 ,65.007  ,1,1,1
#Sta/Elev= 13
   -20.5   74.26   -15.5   71.26   -10.5   68.26      -6   67.26      -3   66.26
      -2   65.96       0   65.96       2   64.46       3   64.46       5   65.86
       6   65.86     8.5   64.06    18.5   64.06
#Mann= 3 , 0 , 0
   -20.5    .033       0       0    .033       0       5    .033       0
Bank Sta=0,5
XS Rating Curve= 0
Exp/Cntr=.3,.1

Type RM Length L Ch R = 1 ,65.006  ,6,6,6
#Sta/Elev= 15
   -20.5   74.26   -15.5   71.26   -10.5   68.26      -6   67.26      -3   66.26
      -2   65.96       0   65.96       2   64.46       2   62.96       3   62.96
       3   64.46       5   65.86       6   65.86     8.5   64.06    18.5   64.06
#Mann= 3 , 0 , 0
   -20.5    .033       0       0    .033       0       5    .033       0
Bank Sta=0,5
XS Rating Curve= 0
Exp/Cntr=.3,.1

Type RM Length L Ch R = 1 ,65      ,22,22,22
#Sta/Elev= 12
   -20.7   74.04   -17.7   72.34   -14.7   70.64   -11.7   68.94    -6.7   67.94
      -4   66.54      -2   65.54       0   65.54       2   62.94       3   62.94
       5   65.44      15   65.44
#Mann= 3 , 0 , 0
   -20.7    .033       0       0    .033       0       5    .033       0
Bank Sta=0,5
XS Rating Curve= 0
Exp/Cntr=.3,.1

Type RM Length L Ch R = 1 ,64.028  ,1,1,1
#Sta/Elev= 12
   -20.7   72.67   -17.7   70.97   -14.7   69.27   -11.7   67.57    -6.7   66.57
      -4   65.17      -2   64.17       0   64.17       2   62.77       3   62.77
       5   64.07      15   64.07
#Mann= 3 , 0 , 0
   -20.7    .033       0       0    .033       0       5    .033       0
Bank Sta=0,5
XS Rating Curve= 0
Exp/Cntr=.3,.1

Type RM Length L Ch R = 1 ,64.027  ,26,26,26
#Sta/Elev= 14
   -20.7   72.67   -17.7   70.97   -14.7   69.27   -11.7   67.57    -6.7   66.57
      -4   65.17      -2   64.17       0   64.17       2   62.77       2   61.57
       3   61.57       3   62.77       5   64.07      15   64.07
#Mann= 3 , 0 , 0
   -20.7    .033       0       0    .033       0       5    .033       0
Bank Sta=0,5
XS Rating Curve= 0
Exp/Cntr=.3,.1

Type RM Length L Ch R = 1 ,64.001  ,1,1,1
#Sta/Elev= 11
   -15.4   65.68   -10.4   64.68    -5.4   63.68    -3.4   62.88       0   62.88
       2   61.28       3   61.28       5   62.78     5.7   62.78     6.1   62.38
    16.1   62.38
#Mann= 3 , 0 , 0
   -15.4    .033       0       0    .033       0       5    .033       0
Bank Sta=0,5
XS Rating Curve= 0
Exp/Cntr=.3,.1

Type RM Length L Ch R = 1 ,64      ,35,35,35
#Sta/Elev= 13
   -15.4   65.68   -10.4   64.68    -5.4   63.68    -3.4   62.88       0   62.88
       2   61.28       2   60.28       3   60.28       3   61.28       5   62.78
     5.7   62.78     6.1   62.38    16.1   62.38
#Mann= 3 , 0 , 0
   -15.4    .033       0       0    .033       0       5    .033       0
Bank Sta=0,5
XS Rating Curve= 0
Exp/Cntr=.3,.1

Type RM Length L Ch R = 1 ,63.015  ,1,1,1
#Sta/Elev= 11
    -8.5   63.98    -6.5   62.98    -4.5   61.98    -2.5   60.98       0   60.98
       2   59.78       3   59.78     4.8   60.98     5.4   60.98     8.6   58.98
    18.6   58.98
#Mann= 3 , 0 , 0
    -8.5    .033       0       0    .033       0     4.8    .033       0
Bank Sta=0,4.8
XS Rating Curve= 0
Exp/Cntr=.3,.1

Type RM Length L Ch R = 1 ,63.014  ,14,14,14
#Sta/Elev= 13
    -8.5   63.98    -6.5   62.98    -4.5   61.98    -2.5   60.98       0   60.98
       2   59.78       2   58.28       3   58.28       3   59.78     4.8   60.98
     5.4   60.98     8.6   58.98    18.6   58.98
#Mann= 3 , 0 , 0
    -8.5    .033       0       0    .033       0     4.8    .033       0
Bank Sta=0,4.8
XS Rating Curve= 0
Exp/Cntr=.3,.1

Type RM Length L Ch R = 1 ,63      ,17,17,17
#Sta/Elev= 12
    -8.5   62.44    -6.5   61.44    -4.5   60.44    -2.5   59.44       0   59.44
       2   58.54       3   58.54     4.8   59.44     5.4   59.44     5.4   59.14
     7.2   57.54    17.2   57.54
#Mann= 3 , 0 , 0
    -8.5    .033       0       0    .033       0     4.8    .033       0
Bank Sta=0,4.8
XS Rating Curve= 0
Exp/Cntr=.3,.1

Type RM Length L Ch R = 1 ,62.033  ,1,1,1
#Sta/Elev= 12
    -8.5   62.33    -6.5   61.33    -4.5   60.33    -2.5   59.33       0   59.33
       2   58.13       3   58.13     4.8   59.33     5.4   59.33     5.4   59.03
     7.2   57.43    17.2   57.43
#Mann= 3 , 0 , 0
    -8.5    .033       0       0    .033       0     4.8    .033       0
Bank Sta=0,4.8
XS Rating Curve= 0
Exp/Cntr=.3,.1

Type RM Length L Ch R = 1 ,62.032  ,32,32,32
#Sta/Elev= 14
    -8.5   62.33    -6.5   61.33    -4.5   60.33    -2.5   59.33       0   59.33
       2   58.13       2   56.93       3   56.93       3   58.13     4.8   59.33
     5.4   59.33     5.4   59.03     7.2   57.43    17.2   57.43
#Mann= 3 , 0 , 0
    -8.5    .033       0       0    .033       0     4.8    .033       0
Bank Sta=0,4.8
XS Rating Curve= 0
Exp/Cntr=.3,.1

Type RM Length L Ch R = 1 ,62      ,1,1,1
#Sta/Elev= 11
    -9.8    61.4    -7.8    60.4    -5.8    59.4    -3.8    58.4       0    58.4
       2    56.8       3    56.8       5    58.3     5.7    58.3     6.2    57.7
    16.2    57.7
#Mann= 3 , 0 , 0
    -9.8    .033       0       0    .033       0       5    .033       0
Bank Sta=0,5
XS Rating Curve= 0
Exp/Cntr=.3,.1

Type RM Length L Ch R = 1 ,61.049  ,1,1,1
#Sta/Elev= 9
    -9.8   61.18    -7.8   60.18    -5.8   59.18    -3.8   58.18       0   58.18
       2   56.38       3   56.38       5   58.08      15   58.08
#Mann= 3 , 0 , 0
    -9.8    .033       0       0    .033       0       5    .033       0
Bank Sta=0,5
XS Rating Curve= 0
Exp/Cntr=.3,.1

Type RM Length L Ch R = 1 ,61.048  ,48,48,48
#Sta/Elev= 11
    -9.8   61.18    -7.8   60.18    -5.8   59.18    -3.8   58.18       0   58.18
       2   56.38       2   55.18       3   55.18       3   56.38       5   58.08
      15   58.08
#Mann= 3 , 0 , 0
    -9.8    .033       0       0    .033       0       5    .033       0
Bank Sta=0,5
XS Rating Curve= 0
Exp/Cntr=.3,.1

Type RM Length L Ch R = 1 ,61      ,30,30,30
#Sta/Elev= 12
   -11.5    61.9    -6.5    59.4    -1.5    56.9       0    56.9      .6    56.3
     2.2    55.2     4.2    55.2     6.2    56.2     7.2    56.8     7.9    56.8
     8.2    56.4    18.2    56.4
#Mann= 3 , 0 , 0
   -11.5    .033       0       0    .033       0     7.2    .033       0
Bank Sta=0,7.2
XS Rating Curve= 0
Exp/Cntr=.3,.1

Type RM Length L Ch R = 1 ,60.02   ,1,1,1
#Sta/Elev= 12
   -11.5   61.71    -6.5   59.21    -1.5   56.71       0   56.71      .6   56.11
     2.2   54.71     3.2   54.71     5.2   56.01     6.2   56.71     6.9   56.71
     7.2   56.31    17.2   56.31
#Mann= 3 , 0 , 0
   -11.5    .033       0       0    .033       0     6.2    .033       0
Bank Sta=0,6.2
XS Rating Curve= 0
Exp/Cntr=.3,.1

Type RM Length L Ch R = 1 ,60.019  ,19,19,19
#Sta/Elev= 14
   -11.5   61.71    -6.5   59.21    -1.5   56.71       0   56.71      .6   56.11
     2.2   54.71     2.2   53.71     3.2   53.71     3.2   54.71     5.2   56.01
     6.2   56.71     6.9   56.71     7.2   56.31    17.2   56.31
#Mann= 3 , 0 , 0
   -11.5    .033       0       0    .033       0     6.2    .033       0
Bank Sta=0,6.2
XS Rating Curve= 0
Exp/Cntr=.3,.1

Type RM Length L Ch R = 1 ,60      ,12,12,12
#Sta/Elev= 9
    -3.2    57.2       0    55.6      .8    55.1     2.8    53.9     3.6    53.9
     4.5    54.4     6.5    55.6     9.5    55.6    12.5    55.6
#Mann= 3 , 0 , 0
    -3.2    .033       0       0    .033       0     6.5    .033       0
Bank Sta=0,6.5
XS Rating Curve= 0
Exp/Cntr=.3,.1

Type RM Length L Ch R = 1 ,59.038  ,24,24,24
#Sta/Elev= 8
     -10   55.18       0   55.18     1.6   54.18     2.2   53.48     3.4   53.48
     5.6   53.88       7   55.28      17   55.28
#Mann= 3 , 0 , 0
     -10    .033       0       0    .033       0       7    .033       0
Bank Sta=0,7
XS Rating Curve= 0
Exp/Cntr=.3,.1

Type RM Length L Ch R = 1 ,59.014  ,14,14,14
#Sta/Elev= 6
     -10   50.88       0   50.88       0   49.28       2   49.28       2   50.88
      12   50.88
#Mann= 3 , 0 , 0
     -10    .033       0       0    .033       0       2    .033       0
Bank Sta=0,2
XS Rating Curve= 0
Exp/Cntr=.3,.1

Type RM Length L Ch R = 1 ,59      ,50,50,50
#Sta/Elev= 12
   -11.3    51.2    -1.3    51.2     -.7    51.6       0    51.6     2.5    50.4
     4.5    49.3     5.9    49.3     7.9    50.4     8.7    50.8     9.3    50.8
    11.5    49.2    21.5    49.2
#Mann= 3 , 0 , 0
   -11.3    .033       0       0    .033       0     8.7    .033       0
Bank Sta=0,8.7
XS Rating Curve= 0
Exp/Cntr=.3,.1

Type RM Length L Ch R = 1 ,58      ,.5,.5,.5
#Sta/Elev= 12
   -11.3   50.38    -1.3   50.38     -.7   50.78       0   50.78     2.5   49.58
     4.5   48.38     5.9   48.38     7.9   49.58     8.7   49.98     9.3   49.98
    11.5   48.38    21.5   48.38
#Mann= 3 , 0 , 0
   -11.3    .033       0       0    .033       0     8.7    .033       0
Bank Sta=0,8.7
XS Rating Curve= 0
Exp/Cntr=.3,.1

Type RM Length L Ch R = 1 ,57.495  ,.5,.5,.5
#Sta/Elev= 12
   -11.3   50.34    -1.3   50.34     -.7   50.74       0   50.74     2.5   49.34
     4.5   48.14     5.9   48.14     7.9   49.34     8.7   49.94     9.3   49.94
    11.5   48.34    21.5   48.34
#Mann= 3 , 0 , 0
   -11.3    .033       0       0    .033       0     8.7    .033       0
Bank Sta=0,8.7
XS Rating Curve= 0
Exp/Cntr=.3,.1

Type RM Length L Ch R = 1 ,57.049  ,49,49,49
#Sta/Elev= 14
   -11.3   50.34    -1.3   50.34     -.7   50.74       0   50.74     2.5   49.34
     4.5   48.14     4.5   47.14     5.9   47.14     5.9   48.14     7.9   49.34
     8.7   49.94     9.3   49.94    11.5   48.34    21.5   48.34
#Mann= 3 , 0 , 0
   -11.3    .033       0       0    .033       0     8.7    .033       0
Bank Sta=0,8.7
XS Rating Curve= 0
Exp/Cntr=.3,.1

Type RM Length L Ch R = 1 ,57      ,26,26,26
#Sta/Elev= 15
   -19.3   56.27   -14.3   54.27    -9.3   52.27    -6.3   49.77    -3.3   49.77
    -1.7   49.27       0   48.47     1.3   47.87     3.3    46.7     4.7   46.77
     6.7   47.87     7.7   48.47     8.2   48.47     9.6   47.37    19.6   47.37
#Mann= 3 , 0 , 0
   -19.3    .033       0    -3.3    .033       0     7.7    .033       0
Bank Sta=-3.3,7.7
XS Rating Curve= 0
Exp/Cntr=.3,.1

Type RM Length L Ch R = 1 ,56.024  ,1,1,1
#Sta/Elev= 15
   -19.5      56   -14.5      54    -9.5      52    -6.5    49.5    -3.5    49.5
    -1.9      49       0    48.1     1.1    47.6     3.1    46.6     4.5    46.6
     6.5    47.6     7.5    48.1       8    48.1     9.4      47    19.4      47
#Mann= 3 , 0 , 0
   -19.5    .033       0    -3.5    .033       0     7.5    .033       0
Bank Sta=-3.5,7.5
XS Rating Curve= 0
Exp/Cntr=.3,.1

Type RM Length L Ch R = 1 ,56.023  ,23,23,23
#Sta/Elev= 17
   -19.5      56   -14.5      54    -9.5      52    -6.5    49.5    -3.5    49.5
    -1.9      49       0    48.1     1.1    47.6     3.1    46.6     3.1    45.1
     4.5    45.1     4.5    46.6     6.5    47.6     7.5    48.1       8    48.1
     9.4      47    19.4      47
#Mann= 3 , 0 , 0
   -19.5    .033       0    -3.5    .033       0     7.5    .033       0
Bank Sta=-3.5,7.5
XS Rating Curve= 0
Exp/Cntr=.3,.1

Type RM Length L Ch R = 1 ,56      ,42,42,42
#Sta/Elev= 12
     -10   52.64      -6   50.14      -2   47.64       0   46.84       2   46.04
       3   45.24     3.6   45.24     4.3   45.54       6   46.54     6.6   46.54
     7.2   46.14    17.2   46.14
#Mann= 3 , 0 , 0
     -10    .033       0       0    .033       0       6    .033       0
Bank Sta=0,6
XS Rating Curve= 0
Exp/Cntr=.3,.1

Type RM Length L Ch R = 1 ,55.008  ,1,1,1
#Sta/Elev= 14
     -14   53.53     -11   52.33      -8   51.13      -5   49.93      -4   49.23
      -2   47.73       0   46.23     1.6   45.83     3.6   44.33     5.2   44.33
     7.7   46.03     8.3   46.03     8.8   45.63    18.8   45.63
#Mann= 3 , 0 , 0
     -14    .033       0       0    .033       0     7.7    .033       0
Bank Sta=0,7.7
XS Rating Curve= 0
Exp/Cntr=.3,.1

Type RM Length L Ch R = 1 ,55.007  ,7,7,7
#Sta/Elev= 16
     -14   53.53     -11   52.33      -8   51.13      -5   49.93      -4   49.23
      -2   47.73       0   46.23     1.6   45.83     3.6   44.33     3.6   43.33
     5.2   43.33     5.2   44.33     7.7   46.03     8.3   46.03     8.8   45.63
    18.8   45.63
#Mann= 3 , 0 , 0
     -14    .033       0       0    .033       0     7.7    .033       0
Bank Sta=0,7.7
XS Rating Curve= 0
Exp/Cntr=.3,.1

Type RM Length L Ch R = 1 ,55      ,50,50,50
#Sta/Elev= 17
   -14.7   48.04    -4.7   48.04    -4.1   48.44    -3.3   48.44    -1.3   46.94
       0   45.94      .7   45.44       2   45.14     3.3   44.14     4.5   44.14
     5.2   44.04       6   44.04     7.6   45.24     9.6   45.94      10   45.94
    10.2   45.74    20.2   45.74
#Mann= 3 , 0 , 0
   -14.7    .033       0    -3.3    .033       0     9.6    .033       0
Bank Sta=-3.3,9.6
XS Rating Curve= 0
Exp/Cntr=.3,.1

Type RM Length L Ch R = 1 ,54      ,50,50,50
#Sta/Elev= 17
   -14.6   47.21    -4.6   47.21      -4   47.61    -3.2   47.61    -1.2   46.11
       0   45.21      .8   44.61     2.1   44.31     3.4   43.31     4.6   43.31
     5.3   43.21     6.1   43.21     7.7   44.41     9.7   45.21    10.1   45.21
    10.3   45.01    20.3   45.01
#Mann= 3 , 0 , 0
   -14.6    .033       0    -3.2    .033       0     9.7    .033       0
Bank Sta=-3.2,9.7
XS Rating Curve= 0
Exp/Cntr=.3,.1

Type RM Length L Ch R = 1 ,53      ,50,50,50
#Sta/Elev= 9
     -10   44.34       0   44.34     2.3   42.74     5.8   42.74     6.3   43.44
     7.5   44.24     8.3   44.24       9   43.64      19   43.64
#Mann= 3 , 0 , 0
     -10    .033       0       0    .033       0     7.5    .033       0
Bank Sta=0,7.5
XS Rating Curve= 0
Exp/Cntr=.3,.1

Type RM Length L Ch R = 1 ,52      ,11,11,11
#Sta/Elev= 9
     -10   44.17       0   44.17     2.8   42.67     6.3   42.67     6.8   43.27
       8   44.07     8.8   44.07     9.5   43.47    19.5   43.47
#Mann= 3 , 0 , 0
     -10    .033       0       0    .033       0       8    .033       0
Bank Sta=0,8
XS Rating Curve= 0
Exp/Cntr=.3,.1

Type RM Length L Ch R = 1 ,51.039  ,39,39,39
#Sta/Elev= 11
   -15.7   43.95    -5.7   43.95    -4.5   44.75       0   44.75       3   42.95
     4.7   42.95     5.2   42.65     6.7   42.65     7.7   43.65     8.5   44.45
    18.5   44.45
#Mann= 3 , 0 , 0
   -15.7    .033       0       0    .033       0     8.5    .033       0
Bank Sta=0,8.5
XS Rating Curve= 0
Exp/Cntr=.3,.1

Type RM Length L Ch R = 1 ,51      ,50,50,50
#Sta/Elev= 6
     -10   44.54       0   44.54     1.2   42.34     3.6   42.34     3.9   44.24
    13.9   44.24
#Mann= 3 , 0 , 0
     -10    .033       0       0    .033       0     3.9    .033       0
Bank Sta=0,3.9
XS Rating Curve= 0
Exp/Cntr=.3,.1

Type RM Length L Ch R = 1 ,50      ,50,50,50
#Sta/Elev= 6
     -10   44.28       0   44.28     1.2   42.08     3.6   42.08     3.9   43.98
    13.9   43.98
#Mann= 3 , 0 , 0
     -10    .033       0       0    .033       0     3.9    .033       0
Bank Sta=0,3.9
XS Rating Curve= 0
Exp/Cntr=.3,.1

Type RM Length L Ch R = 1 ,49      ,8,8,8
#Sta/Elev= 6
     -10    44.2       0    44.2     1.2    42.6     3.6    42.6     3.9    43.9
    13.9    43.9
#Mann= 3 , 0 , 0
     -10    .033       0       0    .033       0     3.9    .033       0
Bank Sta=0,3.9
XS Rating Curve= 0
Exp/Cntr=.3,.1

Type RM Length L Ch R = 1 ,48.042  ,42,42,42
#Sta/Elev= 6
     -10   44.19       0   44.19     1.2   42.69     3.6   42.69     3.9   43.89
    13.9   43.89
#Mann= 3 , 0 , 0
     -10    .033       0       0    .033       0     3.9    .033       0
Bank Sta=0,3.9
XS Rating Curve= 0
Exp/Cntr=.3,.1

Type RM Length L Ch R = 1 ,48      ,25,25,25
#Sta/Elev= 10
     -10   44.48       0   44.48       0   42.28      .9   41.98     4.5   41.98
     4.8   42.28     5.8   42.68     5.8   42.68     5.8   44.58    15.8   44.58
#Mann= 3 , 0 , 0
     -10    .033       0       0    .033       0     5.8    .033       0
Bank Sta=0,5.8
XS Rating Curve= 0
Exp/Cntr=.3,.1

Type RM Length L Ch R = 1 ,47.025  ,1,1,1
#Sta/Elev= 16
   -13.2   41.62    -3.2   41.62    -1.4   42.92       0   42.92     1.4   41.72
       2   41.72     2.3   41.42     2.7   41.42     3.2   41.72     4.2   41.72
     5.8   42.62     7.8   43.52     8.7   43.72    11.7   43.72    12.9   42.82
    22.9   42.82
#Mann= 3 , 0 , 0
   -13.2    .033       0       0    .033       0     8.7    .033       0
Bank Sta=0,8.7
XS Rating Curve= 0
Exp/Cntr=.3,.1

Type RM Length L Ch R = 1 ,47.024  ,24,24,24
#Sta/Elev= 18
   -13.2   41.62    -3.2   41.62    -1.4   42.92       0   42.92     1.4   41.72
       2   41.72     2.3   41.42     2.3   39.92     2.7   39.92     2.7   41.42
     3.2   41.72     4.2   41.72     5.8   42.62     7.8   43.52     8.7   43.72
    11.7   43.72    12.9   42.82    22.9   42.82
#Mann= 3 , 0 , 0
   -13.2    .033       0       0    .033       0     8.7    .033       0
Bank Sta=0,8.7
XS Rating Curve= 0
Exp/Cntr=.3,.1

Type RM Length L Ch R = 1 ,47      ,46,46,46
#Sta/Elev= 11
   -11.1   42.81    -1.1   42.81     -.6   43.21       0   43.21     1.4   42.51
     3.8   39.81     5.4   39.81     7.2   42.21     7.4   42.21    11.4   43.71
    21.4   43.71
#Mann= 3 , 0 , 0
   -11.1    .033       0       0    .033       0    11.4    .033       0
Bank Sta=0,11.4
XS Rating Curve= 0
Exp/Cntr=.3,.1

Type RM Length L Ch R = 1 ,46.004  ,1,1,1
#Sta/Elev= 11
   -11.1   42.21    -1.1   42.21     -.6   42.61       0   42.61     1.4   41.91
     3.8   39.41     5.4   39.41     7.2   41.61     7.4   41.61    11.4   43.11
    21.4   43.11
#Mann= 3 , 0 , 0
   -11.1    .033       0       0    .033       0    11.4    .033       0
Bank Sta=0,11.4
XS Rating Curve= 0
Exp/Cntr=.3,.1

Type RM Length L Ch R = 1 ,46.003  ,3,3,3
#Sta/Elev= 13
   -11.1   42.21    -1.1   42.21     -.6   42.61       0   42.61     1.4   41.91
     3.8   39.41     3.8   38.21     5.4   38.21     5.4   39.41     7.2   41.61
     7.4   41.61    11.4   43.11    21.4   43.11
#Mann= 3 , 0 , 0
   -11.1    .033       0       0    .033       0    11.4    .033       0
Bank Sta=0,11.4
XS Rating Curve= 0
Exp/Cntr=.3,.1

Type RM Length L Ch R = 1 ,46      ,50,50,50
#Sta/Elev= 11
   -11.1   41.44    -1.1   41.44     -.6   41.84       0   41.84     1.4   39.84
     3.8   38.24     5.4   38.24     7.2   40.84     7.4   40.84    11.4   42.34
    21.4   42.34
#Mann= 3 , 0 , 0
   -11.1    .033       0       0    .033       0    11.4    .033       0
Bank Sta=0,11.4
XS Rating Curve= 0
Exp/Cntr=.3,.1

Type RM Length L Ch R = 1 ,45      ,50,50,50
#Sta/Elev= 13
   -11.6   39.21    -1.6   39.21    -1.1   39.21     -.3   39.71       0   39.71
     1.6   38.41     2.1   37.61     3.8   37.61     4.3   38.31     6.3   39.91
     7.3   39.91     8.3   38.91    18.3   38.91
#Mann= 3 , 0 , 0
   -11.6    .033       0       0    .033       0     6.3    .033       0
Bank Sta=0,6.3
XS Rating Curve= 0
Exp/Cntr=.3,.1

Type RM Length L Ch R = 1 ,44      ,23,23,23
#Sta/Elev= 13
   -11.6   39.03    -1.6   39.03    -1.1   39.03     -.3   39.53       0   39.53
     1.6   38.33     2.1   37.73     3.8   37.73     4.3   38.23     6.3   39.53
     7.3   39.53     8.3   38.53    18.3   38.53
#Mann= 3 , 0 , 0
   -11.6    .033       0       0    .033       0     6.3    .033       0
Bank Sta=0,6.3
XS Rating Curve= 0
Exp/Cntr=.3,.1

Type RM Length L Ch R = 1 ,42.027  ,1,1,1
#Sta/Elev= 10
   -11.5   38.39    -1.5   38.39      -1   38.69       0   38.69       2   37.29
       4   37.29       6   38.69     6.8   38.69     8.8   37.09    18.8   37.09
#Mann= 3 , 0 , 0
   -11.5    .033       0       0    .033       0       6    .033       0
Bank Sta=0,6
XS Rating Curve= 0
Exp/Cntr=.3,.1

Type RM Length L Ch R = 1 ,42.026  ,26,26,26
#Sta/Elev= 12
   -11.5   38.39    -1.5   38.39      -1   38.69       0   38.69       2   37.29
       2   36.29       4   36.29       4   37.29       6   38.69     6.8   38.69
     8.8   37.09    18.8   37.09
#Mann= 3 , 0 , 0
   -11.5    .033       0       0    .033       0       6    .033       0
Bank Sta=0,6
XS Rating Curve= 0
Exp/Cntr=.3,.1

Type RM Length L Ch R = 1 ,42      ,50,50,50
#Sta/Elev= 19
   -23.5   43.03   -13.5   43.03   -11.3   41.83    -9.3   40.53    -7.3   39.03
    -6.8   39.03    -5.4   40.23    -2.6   40.23    -1.6   39.13       0   38.23
     1.8   37.43     3.4   37.13     4.4   37.03     4.9   36.53     5.7   36.53
     8.2   37.93     9.2   37.93    10.4   36.93    20.4   36.93
#Mann= 3 , 0 , 0
   -23.5    .033       0    -2.6    .033       0     8.2    .033       0
Bank Sta=-2.6,8.2
XS Rating Curve= 0
Exp/Cntr=.3,.1

Type RM Length L Ch R = 1 ,41      ,41,41,41
#Sta/Elev= 11
      -6      39      -4    38.8      -2    38.4       0    38.1       0    36.6
      .6      36       4      36     4.3    36.3     5.5    37.1     5.5    37.8
    15.5    37.8
#Mann= 3 , 0 , 0
      -6    .033       0       0    .033       0     5.5    .033       0
Bank Sta=0,5.5
XS Rating Curve= 0
Exp/Cntr=.3,.1

Type RM Length L Ch R = 1 ,40.009  ,8,8,8
#Sta/Elev= 11
      -6   39.02      -4   38.72      -2   38.42       0   38.12       0   36.62
      .6   35.92       4   35.92     4.3   36.32     5.5   37.22     5.5   38.12
    15.5   38.12
#Mann= 3 , 0 , 0
      -6    .033       0       0    .033       0     5.5    .033       0
Bank Sta=0,5.5
XS Rating Curve= 0
Exp/Cntr=.3,.1

Type RM Length L Ch R = 1 ,40.001  ,1,1,1
#Sta/Elev= 14
   -15.1   39.49    -5.1   39.49    -3.7   38.79    -2.1   37.29    -1.6   37.29
     -.6   38.09       0   38.09     1.6   37.09       3   36.09     6.2   36.09
     8.2   37.29       9   37.29    10.8   35.89    20.8   35.89
#Mann= 3 , 0 , 0
   -15.1    .033       0       0    .033       0     8.2    .033       0
Bank Sta=0,8.2
XS Rating Curve= 0
Exp/Cntr=.3,.1

Type RM Length L Ch R = 1 ,40      ,50,50,50
#Sta/Elev= 16
   -15.1   39.49    -5.1   39.49    -3.7   38.79    -2.1   37.29    -1.6   37.29
     -.6   38.09       0   38.09     1.6   37.09       3   36.09       3   35.29
     6.2   35.29     6.2   36.09     8.2   37.29       9   37.29    10.8   35.89
    20.8   35.89
#Mann= 3 , 0 , 0
   -15.1    .033       0       0    .033       0     8.2    .033       0
Bank Sta=0,8.2
XS Rating Curve= 0
Exp/Cntr=.3,.1

Type RM Length L Ch R = 1 ,39      ,29,29,29
#Sta/Elev= 10
   -14.5   38.24    -4.5   38.24      -2   36.64       0   36.64     1.6   34.94
     4.4   34.94     6.6   36.64     7.2   36.64     7.8   36.24    17.8   36.24
#Mann= 3 , 0 , 0
   -14.5    .033       0       0    .033       0     6.6    .033       0
Bank Sta=0,6.6
XS Rating Curve= 0
Exp/Cntr=.3,.1

Type RM Length L Ch R = 1 ,38.021  ,1,1,1
#Sta/Elev= 10
   -14.5   37.84    -4.5   37.84      -2   36.24       0   36.24     1.6   35.04
     4.4   35.04     6.6   36.24     7.2   36.24     7.8   35.84    17.8   35.84
#Mann= 3 , 0 , 0
   -14.5    .033       0       0    .033       0     6.6    .033       0
Bank Sta=0,6.6
XS Rating Curve= 0
Exp/Cntr=.3,.1

Type RM Length L Ch R = 1 ,38.02   ,20,20,20
#Sta/Elev= 12
   -14.5   37.84    -4.5   37.84      -2   36.24       0   36.24     1.6   35.04
     1.6   34.04     4.4   34.04     4.4   35.04     6.6   36.24     7.2   36.24
     7.8   35.84    17.8   35.84
#Mann= 3 , 0 , 0
   -14.5    .033       0       0    .033       0     6.6    .033       0
Bank Sta=0,6.6
XS Rating Curve= 0
Exp/Cntr=.3,.1

Type RM Length L Ch R = 1 ,38      ,50,50,50
#Sta/Elev= 13
   -15.2    37.4    -5.2    37.4    -4.2    37.1    -1.7    35.4       0    35.4
       2    33.9     3.2    33.9     3.6    34.2     4.1    34.3     6.1    35.6
     6.9    35.6     7.5    35.1    17.5    35.1
#Mann= 3 , 0 , 0
   -15.2    .033       0       0    .033       0     6.1    .033       0
Bank Sta=0,6.1
XS Rating Curve= 0
Exp/Cntr=.3,.1

Type RM Length L Ch R = 1 ,37      ,36,36,36
#Sta/Elev= 13
   -15.2   37.29    -5.2   37.29    -4.2   36.99    -1.7   35.29       0   35.29
       2   33.79     3.2   33.79     3.6   34.09     4.1   34.19     6.1   35.39
     6.9   35.39     7.5   34.89    17.5   34.89
#Mann= 3 , 0 , 0
   -15.2    .033       0       0    .033       0     6.1    .033       0
Bank Sta=0,6.1
XS Rating Curve= 0
Exp/Cntr=.3,.1

Type RM Length L Ch R = 1 ,36.014  ,14,14,14
#Sta/Elev= 6
     -10   36.15       0   36.15       0   33.65     2.7   33.65     2.7   36.15
    12.7   36.15
#Mann= 3 , 0 , 0
     -10    .033       0       0    .033       0     2.7    .033       0
Bank Sta=0,2.7
XS Rating Curve= 0
Exp/Cntr=.3,.1

Type RM Length L Ch R = 1 ,36      ,50,50,50
#Sta/Elev= 6
     -10   35.74       0   35.74       0   33.24     2.7   33.24     2.7   35.74
    12.7   35.74
#Mann= 3 , 0 , 0
     -10    .033       0       0    .033       0     2.7    .033       0
Bank Sta=0,2.7
XS Rating Curve= 0
Exp/Cntr=.3,.1

Type RM Length L Ch R = 1 ,35      ,50,50,50
#Sta/Elev= 15
   -11.6   33.99    -1.6   33.99     -.6   34.69       0   34.69     1.6   33.59
     2.6   33.59     3.4   33.09     4.2   33.09     4.9   33.49     5.7   33.89
     7.1   35.19     9.1   35.89    11.4   37.79    12.6   37.79    22.6   37.79
#Mann= 3 , 0 , 0
   -11.6    .033       0       0    .033       0    11.4    .033       0
Bank Sta=0,11.4
XS Rating Curve= 0
Exp/Cntr=.3,.1

Type RM Length L Ch R = 1 ,34      ,37,37,37
#Sta/Elev= 15
   -11.6   33.65    -1.6   33.65     -.6   34.35       0   34.35     1.6   33.25
     2.6   33.25     3.4   32.75     4.2   32.75     4.9   33.15     5.7   33.55
     7.1   34.85     9.1   35.55    11.4   37.45    12.6   37.45    22.6   37.45
#Mann= 3 , 0 , 0
   -11.6    .033       0       0    .033       0    11.4    .033       0
Bank Sta=0,11.4
XS Rating Curve= 0
Exp/Cntr=.3,.1

Type RM Length L Ch R = 1 ,33.013  ,13,13,13
#Sta/Elev= 14
   -12.1   33.76    -2.1   33.76     -.7   34.56       0   34.56      .7   34.06
      .9   34.06     2.4   32.76     5.9   32.76     7.4   34.16     7.6   34.16
     8.8   35.26    11.2   35.26    12.3   34.26    22.3   34.26
#Mann= 3 , 0 , 0
   -12.1    .033       0       0    .033       0     8.8    .033       0
Bank Sta=0,8.8
XS Rating Curve= 0
Exp/Cntr=.3,.1

Type RM Length L Ch R = 1 ,32      ,14,14,14
#Sta/Elev= 15
   -11.3    34.2    -1.3    34.2     -.5    34.7       0    34.7     1.4    33.7
     2.4    32.6     3.2    32.4     3.7    31.9     4.5    31.9     5.5    32.4
     6.8    32.8     9.2    34.2      10    34.2    11.1    33.4    21.1    33.4
#Mann= 3 , 0 , 0
   -11.3    .033       0       0    .033       0     9.2    .033       0
Bank Sta=0,9.2
XS Rating Curve= 0
Exp/Cntr=.3,.1

Type RM Length L Ch R = 1 ,31.036  ,1,1,1
#Sta/Elev= 12
   -11.4   33.75    -1.4   33.75     -.6   34.45       0   34.45     1.2   33.65
     2.8   32.25     5.4   32.25     7.2   33.45     8.8   34.25    9.47   34.25
    10.4   33.45    20.4   33.45
#Mann= 3 , 0 , 0
   -11.4    .033       0       0    .033       0     8.8    .033       0
Bank Sta=0,8.8
XS Rating Curve= 0
Exp/Cntr=.3,.1

Type RM Length L Ch R = 1 ,31.035  ,35,35,35
#Sta/Elev= 14
   -11.4   33.75    -1.4   33.75     -.6   34.45       0   34.45     1.2   33.65
     2.8   32.25     2.8   31.55     5.4   31.55     5.4   32.25     7.2   33.45
     8.8   34.25     9.4   34.25    10.4   33.45    20.4   33.45
#Mann= 3 , 0 , 0
   -11.4    .033       0       0    .033       0     8.8    .033       0
Bank Sta=0,8.8
XS Rating Curve= 0
Exp/Cntr=.3,.1

Type RM Length L Ch R = 1 ,31      ,50,50,50
#Sta/Elev= 12
   -11.2   32.84    -1.2   32.84     -.6   33.34       0   33.34     2.3   31.44
     3.3   31.44     3.7   32.04     4.2   32.04     5.9   33.84     6.6   33.84
     7.1   33.54    17.1   33.54
#Mann= 3 , 0 , 0
   -11.2    .033       0       0    .033       0     5.9    .033       0
Bank Sta=0,5.9
XS Rating Curve= 0
Exp/Cntr=.3,.1

Type RM Length L Ch R = 1 ,30      ,50,50,50
#Sta/Elev= 12
   -11.2   32.05    -1.2   32.05     -.6   32.55       0   32.55     2.3   30.95
     3.3   30.95     3.7   31.25     4.2   31.25     5.9   32.65     6.6   32.65
     7.1   32.35    17.1   32.35
#Mann= 3 , 0 , 0
   -11.2    .033       0       0    .033       0     5.9    .033       0
Bank Sta=0,5.9
XS Rating Curve= 0
Exp/Cntr=.3,.1

Type RM Length L Ch R = 1 ,29      ,50,50,50
#Sta/Elev= 13
   -12.1    31.2    -2.1    31.2      -1    31.7       0    31.7     1.6    30.3
     2.2    30.1       3    30.1     3.9    30.4     5.1    30.5     7.1    32.3
     7.7    32.3     9.5    30.8    19.5    30.8
#Mann= 3 , 0 , 0
   -12.1    .033       0       0    .033       0     7.1    .033       0
Bank Sta=0,7.1
XS Rating Curve= 0
Exp/Cntr=.3,.1

Type RM Length L Ch R = 1 ,28      ,50,50,50
#Sta/Elev= 13
   -12.1   31.21    -2.1   31.21      -1   31.71       0   31.71     1.6   30.51
     2.2   30.11       3   30.11     3.9   30.51     5.1   30.61     7.1   32.31
     7.7   32.31     9.5   30.81    19.5   30.81
#Mann= 3 , 0 , 0
   -12.1    .033       0       0    .033       0     7.1    .033       0
Bank Sta=0,7.1
XS Rating Curve= 0
Exp/Cntr=.3,.1

Type RM Length L Ch R = 1 ,27      ,50,50,50
#Sta/Elev= 13
   -12.1   30.39    -2.1   30.39      -1   30.89       0   30.89     1.6   29.79
     2.2   29.49       3   29.49     3.9   29.89     5.1   29.99     7.1   31.59
     7.7   31.59     9.5   30.09    19.5   30.09
#Mann= 3 , 0 , 0
   -12.1    .033       0       0    .033       0     7.1    .033       0
Bank Sta=0,7.1
XS Rating Curve= 0
Exp/Cntr=.3,.1

Type RM Length L Ch R = 1 ,26      ,50,50,50
#Sta/Elev= 20
   -12.5   30.04    -2.6   30.04    -1.4   30.74       0   30.74       1   30.04
       1   29.54     1.4   29.54     1.4   29.34     2.4   29.34     2.4   30.14
     2.7   30.14     2.7   29.34     3.9   29.34     3.9   30.34     4.5   30.74
     5.2   30.74     5.5   31.04       7   31.04     8.7   29.84    18.7   29.84
#Mann= 3 , 0 , 0
   -12.5    .033       0       0    .033       0     5.5    .033       0
Bank Sta=0,5.5
XS Rating Curve= 0
Exp/Cntr=.3,.1

Type RM Length L Ch R = 1 ,25      ,50,50,50
#Sta/Elev= 14
   -12.5   29.94    -2.5   29.94      -1   30.74       0   30.74     1.8   29.34
     2.6   28.84     3.1   28.34       4   28.24       5   28.24     5.2   29.14
     7.7   30.74     8.3   30.74     9.3   29.84    19.3   29.84
#Mann= 3 , 0 , 0
   -12.5    .033       0       0    .033       0     7.7    .033       0
Bank Sta=0,7.7
XS Rating Curve= 0
Exp/Cntr=.3,.1

Type RM Length L Ch R = 1 ,24      ,13,13,13
#Sta/Elev= 14
   -12.5   29.57    -2.5   29.57      -1   30.37       0   30.37     1.8   28.97
     2.6   28.47     3.1   27.97       4   27.77       5   27.77     5.2   28.67
     7.7   30.37     8.3   30.37     9.3   29.47    19.3   29.47
#Mann= 3 , 0 , 0
   -12.5    .033       0       0    .033       0     7.7    .033       0
Bank Sta=0,7.7
XS Rating Curve= 0
Exp/Cntr=.3,.1

Type RM Length L Ch R = 1 ,23.037  ,37,37,37
#Sta/Elev= 14
     -13    29.9      -3    29.9      -3    30.9       0    30.9       0    28.7
       2    28.7     2.5      28     4.5      28     6.3    30.5     8.3    30.5
     9.5    30.8     9.7    30.8     9.9    30.6    19.9    30.6
#Mann= 3 , 0 , 0
     -13    .033       0       0    .033       0     9.5    .033       0
Bank Sta=0,9.5
XS Rating Curve= 0
Exp/Cntr=.3,.1

Type RM Length L Ch R = 1 ,23      ,50,50,50
#Sta/Elev= 14
   -12.2   29.01    -2.2   29.01     -.8   30.01       0   30.01     1.8   28.61
     2.3   28.51     4.8   27.81     7.3   27.81     7.7   28.71     8.7   28.81
    10.4   29.91    11.3   29.91    12.3   29.01    22.3   29.01
#Mann= 3 , 0 , 0
   -12.2    .033       0       0    .033       0    10.4    .033       0
Bank Sta=0,10.4
XS Rating Curve= 0
Exp/Cntr=.3,.1

Type RM Length L Ch R = 1 ,22      ,40,40,40
#Sta/Elev= 14
   -12.2   28.79    -2.2   28.79     -.8   29.79       0   29.79     1.8   28.39
     2.3   28.29     2.8   27.59     5.3   27.59     5.7   28.49     6.7   28.59
     8.4   29.69     9.3   29.69    10.3   28.79    20.3   28.79
#Mann= 3 , 0 , 0
   -12.2    .033       0       0    .033       0     8.4    .033       0
Bank Sta=0,8.4
XS Rating Curve= 0
Exp/Cntr=.3,.1

Type RM Length L Ch R = 1 ,21.01   ,10,10,10
#Sta/Elev= 16
     -12   28.53      -2   28.53    -1.2   29.23       0   29.23     1.8   28.33
     1.8   27.73     3.2   27.73     3.2   28.13     4.4   28.13     4.4   28.33
     4.8   28.33     4.8   28.53       7   29.53     7.8   29.53     9.1   28.33
    19.1   28.33
#Mann= 3 , 0 , 0
     -12    .033       0       0    .033       0       7    .033       0
Bank Sta=0,7
XS Rating Curve= 0
Exp/Cntr=.3,.1

Type RM Length L Ch R = 1 ,21      ,50,50,50
#Sta/Elev= 13
   -11.9   28.81    -1.9   28.81     -.7   29.61       0   29.61     1.2   28.61
     3.2   27.01     4.2   27.01     4.9   27.31     5.4   27.71     8.4   29.51
     9.1   29.51      10   28.61      20   28.61
#Mann= 3 , 0 , 0
   -11.9    .033       0       0    .033       0     8.4    .033       0
Bank Sta=0,8.4
XS Rating Curve= 0
Exp/Cntr=.3,.1

Type RM Length L Ch R = 1 ,20      ,50,50,50
#Sta/Elev= 13
   -11.9   28.47    -1.9   28.47     -.7   29.27       0   29.27     1.2   28.27
     3.2   26.77     4.2   26.77     4.9   27.07     5.4   27.47     8.4   29.17
     9.1   29.17      10   28.27      20   28.27
#Mann= 3 , 0 , 0
   -11.9    .033       0       0    .033       0     8.4    .033       0
Bank Sta=0,8.4
XS Rating Curve= 0
Exp/Cntr=.3,.1

Type RM Length L Ch R = 1 ,19      ,12,12,12
#Sta/Elev= 13
     -13    27.9      -3    27.9      -2    28.7       0    28.7       2    27.3
       3    26.4     5.4    26.4     7.2    26.8     8.6    27.2     9.6    29.2
    11.1    29.2    12.8    28.6    22.8    28.6
#Mann= 3 , 0 , 0
     -13    .033       0       0    .033       0     9.6    .033       0
Bank Sta=0,9.6
XS Rating Curve= 0
Exp/Cntr=.3,.1

Type RM Length L Ch R = 1 ,18.038  ,38,38,38
#Sta/Elev= 13
     -13   27.75      -3   27.75      -2   28.55       0   28.55       2   27.15
       3   26.35     5.4   26.35     7.2   26.65     8.6   26.95     9.6   28.75
    11.1   28.75    12.8   28.15    22.8   28.15
#Mann= 3 , 0 , 0
     -13    .033       0       0    .033       0     9.6    .033       0
Bank Sta=0,9.6
XS Rating Curve= 0
Exp/Cntr=.3,.1

Type RM Length L Ch R = 1 ,18      ,50,50,50
#Sta/Elev= 12
   -12.8   27.79    -2.8   27.79      -2   28.29       0   28.29     1.2   27.49
     2.2   26.29     5.4   26.29     6.2   27.59     7.8   28.69     9.1   28.69
     9.5   28.19    19.5   28.19
#Mann= 3 , 0 , 0
   -12.8    .033       0       0    .033       0     7.8    .033       0
Bank Sta=0,7.8
XS Rating Curve= 0
Exp/Cntr=.3,.1

Type RM Length L Ch R = 1 ,17      ,50,50,50
#Sta/Elev= 14
   -12.7   27.65    -2.7   27.65      -2   28.15       0   28.15     1.2   27.45
     1.4   26.45       2   26.05     5.4   26.05     5.8   26.45     6.3   27.35
     7.5   28.25     8.7   28.25     9.6   27.45    19.6   27.45
#Mann= 3 , 0 , 0
   -12.7    .033       0       0    .033       0     7.5    .033       0
Bank Sta=0,7.5
XS Rating Curve= 0
Exp/Cntr=.3,.1

Type RM Length L Ch R = 1 ,16      ,37,37,37
#Sta/Elev= 14
   -12.7   27.45    -2.7   27.45      -2   27.95       0   27.95     1.2   27.25
     1.4   26.25       2   25.95     5.4   25.95     5.8   26.35     6.3   27.25
     7.5   28.05     8.7   28.05     9.6   27.25    19.6   27.25
#Mann= 3 , 0 , 0
   -12.7    .033       0       0    .033       0     7.5    .033       0
Bank Sta=0,7.5
XS Rating Curve= 0
Exp/Cntr=.3,.1

Type RM Length L Ch R = 1 ,15.013  ,13,13,13
#Sta/Elev= 19
   -13.6   26.98    -3.6   26.98      -2   27.98       0   27.98       1   26.88
       1   26.48     2.2   26.48     2.2   25.98     3.2   25.98     3.2   26.58
       5   26.58       5   26.98     5.6   26.98       6   27.38     6.4   27.38
     7.6   27.98     8.8   27.98     9.8   27.48    19.8   27.48
#Mann= 3 , 0 , 0
   -13.6    .033       0       0    .033       0     7.6    .033       0
Bank Sta=0,7.6
XS Rating Curve= 0
Exp/Cntr=.3,.1

Type RM Length L Ch R = 1 ,15      ,50,50,50
#Sta/Elev= 13
     -13   27.52      -3   27.52      -2   28.22       0   28.22     1.5   27.22
     2.8   26.82     3.4   25.82     6.4   25.82     6.7   26.42     9.9   27.82
    10.3   27.82    10.9   27.32    20.9   27.32
#Mann= 3 , 0 , 0
     -13    .033       0       0    .033       0     9.9    .033       0
Bank Sta=0,9.9
XS Rating Curve= 0
Exp/Cntr=.3,.1

Type RM Length L Ch R = 1 ,14      ,50,50,50
#Sta/Elev= 13
     -13    27.2      -3    27.2      -2    27.9       0    27.9     1.5    26.9
     2.8    26.5     3.4    25.4     6.4    25.4     6.7    26.1     9.9    27.7
    10.3    27.7    10.9    27.2    20.9    27.2
#Mann= 3 , 0 , 0
     -13    .033       0       0    .033       0     9.9    .033       0
Bank Sta=0,9.9
XS Rating Curve= 0
Exp/Cntr=.3,.1

Type RM Length L Ch R = 1 ,13      ,1,1,1
#Sta/Elev= 12
   -15.3   27.07    -5.3   27.07    -5.3   27.67       0   27.67       0   25.67
      .2   25.67      .2   25.37     4.6   25.37     4.6   25.67     4.8   25.67
     5.4   27.47    15.4   27.47
#Mann= 3 , 0 , 0
   -15.3    .033       0       0    .033       0     5.4    .033       0
Bank Sta=0,5.4
XS Rating Curve= 0
Exp/Cntr=.3,.1

Type RM Length L Ch R = 1 ,12.049  ,49,49,49
#Sta/Elev= 12
   -15.3   26.79    -5.3   26.79    -5.3   27.39       0   27.39       0   25.79
      .2   25.79      .2   25.39     4.6   25.39     4.6   25.79     4.8   25.79
     5.4   27.39    15.4   27.39
#Mann= 3 , 0 , 0
   -15.3    .033       0       0    .033       0     5.4    .033       0
Bank Sta=0,5.4
XS Rating Curve= 0
Exp/Cntr=.3,.1

Type RM Length L Ch R = 1 ,12      ,29,29,29
#Sta/Elev= 15
   -13.5   26.16    -3.5   26.16      -3   26.46       0   26.46      .4   24.86
       1   24.86     1.4   24.56     3.2   24.56     3.8   24.76     4.4   25.46
       5   25.56     5.4   26.86       8   26.86     9.1   25.86    19.1   25.86
#Mann= 3 , 0 , 0
   -13.5    .033       0       0    .033       0     5.4    .033       0
Bank Sta=0,5.4
XS Rating Curve= 0
Exp/Cntr=.3,.1

Type RM Length L Ch R = 1 ,11.021  ,21,21,21
#Sta/Elev= 15
   -13.5   25.96    -3.5   25.96      -3   26.26       0   26.26      .4   24.66
       1   24.66     1.4   24.36     3.2   24.36     3.8   24.56     4.4   25.26
       5   25.36     5.4   26.66       8   26.66     9.1   25.66    19.1   25.66
#Mann= 3 , 0 , 0
   -13.5    .033       0       0    .033       0     5.4    .033       0
Bank Sta=0,5.4
XS Rating Curve= 0
Exp/Cntr=.3,.1

Type RM Length L Ch R = 1 ,11      ,50,50,50
#Sta/Elev= 12
   -11.6   25.66    -1.6   25.66     -.6   26.56       0   26.56     1.2   25.86
       2   24.36       6   24.36     6.7   25.36     9.7   26.56    11.7   26.56
    13.5   25.06    23.5   25.06
#Mann= 3 , 0 , 0
   -11.6    .033       0       0    .033       0     9.7    .033       0
Bank Sta=0,9.7
XS Rating Curve= 0
Exp/Cntr=.3,.1

Type RM Length L Ch R = 1 ,10      ,19,19,19
#Sta/Elev= 12
   -11.6   25.53    -1.6   25.53     -.6   26.43       0   26.43     1.2   25.73
       2   24.33       6   24.33     6.7   25.23     9.7   26.33    11.7   26.33
    13.5   24.83    23.5   24.83
#Mann= 3 , 0 , 0
   -11.6    .033       0       0    .033       0     9.7    .033       0
Bank Sta=0,9.7
XS Rating Curve= 0
Exp/Cntr=.3,.1

Type RM Length L Ch R = 1 ,9.031   ,31,31,31
#Sta/Elev= 9
     -10   26.78       0   26.78      .6   25.08     3.1   24.28     5.9   24.28
     6.9   26.38     9.3   26.38      11   24.98      21   24.98
#Mann= 3 , 0 , 0
     -10    .033       0       0    .033       0     6.9    .033       0
Bank Sta=0,6.9
XS Rating Curve= 0
Exp/Cntr=.3,.1

Type RM Length L Ch R = 1 ,9       ,42,42,42
#Sta/Elev= 23
   -13.4   24.82    -3.4   24.82    -1.2   26.22       0   26.22      .4   24.52
     1.8   24.22     2.2   23.82     3.2   23.82     3.4   24.02     4.1   24.02
     4.8   24.72     5.4   24.72     5.8   26.22     6.3   26.22     6.8   25.62
     8.5   25.62    11.1   25.32    11.5   24.92    12.1   24.92    12.9   25.82
    13.4   25.82    13.7   25.62    23.7   25.62
#Mann= 3 , 0 , 0
   -13.4    .033       0       0    .033       0     5.8    .033       0
Bank Sta=0,5.8
XS Rating Curve= 0
Exp/Cntr=.3,.1

Type RM Length L Ch R = 1 ,8.008   ,8,8,8
#Sta/Elev= 23
   -13.4   24.56    -3.4   24.56    -1.2   25.96       0   25.96      .4   24.26
     1.8   23.96     2.2   23.46     3.2   23.46     3.4   23.66     4.1   23.66
     4.8   24.36     5.4   24.36     5.8   25.96     6.3   25.96     6.8   25.36
     8.5   25.36    11.1   25.06    11.5   24.66    12.1   24.66    12.9   25.56
    13.4   25.56    13.7   25.36    23.7   25.36
#Mann= 3 , 0 , 0
   -13.4    .033       0       0    .033       0     5.8    .033       0
Bank Sta=0,5.8
XS Rating Curve= 0
Exp/Cntr=.3,.1

Type RM Length L Ch R = 1 ,8       ,50,50,50
#Sta/Elev= 13
   -11.9   24.65    -1.9   24.65     -.5   25.55       0   25.55       2   23.85
     2.9   23.85     3.7   23.55     5.6   23.55     5.9   24.25     7.7   25.25
     9.9   25.25    10.3   24.95    20.3   24.95
#Mann= 3 , 0 , 0
   -11.9    .033       0       0    .033       0     7.7    .033       0
Bank Sta=0,7.7
XS Rating Curve= 0
Exp/Cntr=.3,.1

Type RM Length L Ch R = 1 ,7       ,50,50,50
#Sta/Elev= 12
   -11.6   24.36    -1.6   24.36     -.4   25.16       0   25.16       2   23.36
     4.5   23.36     5.5   24.36       6   24.86     6.5   25.36     8.3   25.36
     9.3   24.56    19.3   24.56
#Mann= 3 , 0 , 0
   -11.6    .033       0       0    .033       0     6.5    .033       0
Bank Sta=0,6.5
XS Rating Curve= 0
Exp/Cntr=.3,.1

Type RM Length L Ch R = 1 ,6       ,50,50,50
#Sta/Elev= 12
   -11.6   23.95    -1.6   23.95     -.4   24.75       0   24.75       2   23.05
     4.5   23.05     5.5   24.05       6   24.45     6.5   24.85     8.3   24.85
     9.3   24.05    19.3   24.05
#Mann= 3 , 0 , 0
   -11.6    .033       0       0    .033       0     6.5    .033       0
Bank Sta=0,6.5
XS Rating Curve= 0
Exp/Cntr=.3,.1

Type RM Length L Ch R = 1 ,5       ,50,50,50
#Sta/Elev= 12
      -6   28.69      -3   26.99       0   25.29       3   23.59     4.2   22.99
     7.2   22.99     8.1   23.39     9.1   23.69    10.3   24.69    11.9   24.69
    13.2   23.69    23.2   23.69
#Mann= 3 , 0 , 0
      -6    .033       0       0    .033       0    10.3    .033       0
Bank Sta=0,10.3
XS Rating Curve= 0
Exp/Cntr=.3,.1

Type RM Length L Ch R = 1 ,4       ,45,45,45
#Sta/Elev= 12
      -6   28.54      -3   26.84       0   25.14       3   23.44     4.2   22.84
     7.2   22.84     8.1   23.24    9.14   23.54    10.3   24.54    11.9   24.54
    13.2   23.54    23.2   23.54
#Mann= 3 , 0 , 0
      -6    .033       0       0    .033       0    10.3    .033       0
Bank Sta=0,10.3
XS Rating Curve= 0
Exp/Cntr=.3,.1

Type RM Length L Ch R = 1 ,3.005   ,5,5,5
#Sta/Elev= 18
   -10.4   29.27    -8.4   28.07    -6.4   26.87    -4.4   25.67    -2.7   25.67
      -2   25.97       0   25.97       2   24.27     3.2   24.27     3.4   22.67
     5.1   22.77     6.1   22.97     8.1   23.07     8.6   24.47    10.3   25.07
    12.5   25.07    14.2   23.37    24.2   23.37
#Mann= 3 , 0 , 0
   -10.4    .033       0       0    .033       0    10.3    .033       0
Bank Sta=0,10.3
XS Rating Curve= 0
Exp/Cntr=.3,.1

Type RM Length L Ch R = 1 ,3       ,50,50,50
#Sta/Elev= 17
   -10.7   31.85    -5.7   28.85     -.7   25.85       0   24.95      .8   23.85
       2   22.65     5.3   22.65     6.2   23.15     6.5   24.45       7   24.95
     9.5   24.95      11   23.95    12.5   23.95    13.1   24.45    13.7   24.45
      14   24.15      24   24.15
#Mann= 3 , 0 , 0
   -10.7    .033       0       0    .033       0       7    .033       0
Bank Sta=0,7
XS Rating Curve= 0
Exp/Cntr=.3,.1

Type RM Length L Ch R = 1 ,2       ,50,50,50
#Sta/Elev= 17
     -11   31.12      -6   28.12      -1   25.12       0   23.82      .5   23.12
     1.7   22.02       5   22.02     5.9   22.42     6.2   23.52     6.7   23.82
     9.2   23.82    10.7   22.82    12.2   22.82    12.8   23.32    13.4   23.32
    13.7   23.02    23.7   23.02
#Mann= 3 , 0 , 0
     -11    .033       0       0    .033       0     6.7    .033       0
Bank Sta=0,6.7
XS Rating Curve= 0
Exp/Cntr=.3,.1
